HEC-RAS study GLADYFK.prj: GLADYFK

--- GLADYFK.g01 (geometry) --- (continued)

Type RM Length L Ch R = 1 ,139932  ,274.2,276,277.4
XS GIS Cut Line= 2
2338428.49090247665702.3615900542339079.09151095665871.289467345
#Sta/Elev= 30
       0 2853.36     7.9 2851.43    16.2 2846.48    45.1 2835.52    65.8 2829.37
   115.4 2821.89     165 2819.24   177.4 2820.48   181.5 2819.65   193.9 2819.36
     227 2820.12   272.4 2819.84   301.4 2815.89   334.4 2817.31   338.5 2816.92
   342.7 2815.49   350.9 2811.08     364 2808.64   379.3 2808.19   400.5 2808.33
     446 2813.53   466.7 2821.94   479.1 2831.43   487.3 2836.33   536.9 2853.81
   582.4 2867.42   594.8 2869.76   607.2  2874.1     665 2888.73   672.2 2889.56
#Mann= 3 ,-1,0
       0      .1       0     364    .045       0   400.5      .1       0
#XS Ineff= 2 , 0
          332.79 2832.04
Permanent Ineff=
       F       F
Bank Sta=364,400.5
XS Rating Curve= 0 ,0
Exp/Cntr(USF)=0,0
Exp/Cntr=0.3,0.1

Type RM Length L Ch R = 1 ,139656  ,302.9,294,277.2
XS GIS Cut Line= 3
2338256.44191646665896.4263598852338840.93071977666103.806807189
2338895.99030597666119.401359885
#Sta/Elev= 30
       0 2942.61    26.2 2935.12    93.1 2905.39   114.3 2896.76   125.7 2893.35
   148.3 2881.29   169.6 2872.67   182.2 2864.45   200.9 2857.93   216.2 2850.05
   235.3 2842.39   272.9 2830.45   305.3 2823.78   316.8 2822.95   330.8 2818.45
   348.1 2815.56   360.5  2815.3   377.5 2817.47   445.7 2807.78   470.3  2807.7
   480.7 2807.76   487.8 2808.05   500.5 2816.17     509 2818.04     560 2821.29
   572.7  2823.1   585.4 2822.88   598.2 2825.88   610.9 2826.39   677.4 2834.97
#Mann= 3 ,-1,0
       0      .1       0   445.7    .045       0   480.7      .1       0
Bank Sta=445.7,480.7
XS Rating Curve= 0 ,0
Exp/Cntr=0.3,0.1

Type RM Length L Ch R = 1 ,139362  ,246.6,237,223.7
XS GIS Cut Line= 2
2338306.89237738666410.7226692162338927.81646688666182.441753959
#Sta/Elev= 30
       0 2857.61    14.7 2856.48      44 2850.32    69.6 2842.31    99.4 2838.38
     125 2837.86   143.6  2839.9   159.1 2839.56   205.9 2833.77   218.7 2830.54
   231.5 2825.19   254.6 2811.03   265.6 2807.43   271.1 2807.27     304 2807.17
   308.2 2807.22     321 2807.33   340.6 2815.73   350.8 2817.95   376.4 2819.55
   423.3 2819.62   440.3 2820.57   448.9 2822.48   465.9 2818.41   470.2 2818.86
   482.9 2824.95   491.5 2824.19   549.3 2827.43   584.1 2822.81   661.6 2832.21
#Mann= 3 ,-1,0
       0      .1       0   271.1    .045       0   308.2      .1       0
Bank Sta=271.1,308.2
XS Rating Curve= 0 ,0
Exp/Cntr(USF)=0,0
Exp/Cntr=0.3,0.1

Type RM Length L Ch R = 1 ,139125  ,266.6,273.7,279.5
XS GIS Cut Line= 2
2338602.76218955666683.4334929312338933.81782459666206.370516655
#Sta/Elev= 30
       0 2918.23    14.1 2913.73    22.8 2913.12    31.4 2908.25    37.6 2907.02
    79.7 2890.02   100.4 2878.81   109.9 2874.92   134.8 2859.92   148.8 2854.24
   163.4  2845.2   173.2 2840.71   184.9 2832.26   197.5 2828.99   209.6 2821.16
   235.4 2813.68   241.3  2811.1   255.9 2809.57   265.7 2806.72   272.8 2806.38
   299.7 2806.34   311.2 2806.38   325.2 2807.63   339.2 2812.61   377.6 2811.64
   390.7 2812.43   402.2 2815.17   445.8 2816.99   518.8 2828.92   580.7 2835.02
#Mann= 3 ,-1,0
       0      .1       0   272.8    .045       0   311.2      .1       0
Bank Sta=272.8,311.2
XS Rating Curve= 0 ,0
Exp/Cntr=0.3,0.1

Type RM Length L Ch R = 1 ,138851  ,203.9,206.1,208.3
XS GIS Cut Line= 2
 2338709.9020312666784.9294021572339246.13390113666396.623565305
#Sta/Elev= 30
       0 2901.06    26.9 2892.77    52.2 2880.06      61 2877.55    71.9 2870.66
    86.8 2864.42      96 2859.43   101.9 2857.83     116 2850.82     136 2843.13
   173.3 2823.37   187.6  2817.5   210.2  2815.3     225 2816.14   267.8 2811.82
   299.1 2812.33   306.5  2814.4   313.3 2814.43   354.2 2805.78   358.4 2805.75
   393.9 2805.78   405.3 2806.36   416.8 2810.61   436.8 2810.32   465.5 2822.96
     497 2825.84   531.4 2832.52   546.1 2837.75     627 2872.99   662.1 2883.59
#Mann= 3 ,-1,0
       0      .1       0   354.2    .045       0   393.9      .1       0
Bank Sta=354.2,393.9
XS Rating Curve= 0 ,0
Exp/Cntr(USF)=0,0
Exp/Cntr=0.3,0.1

Type RM Length L Ch R = 1 ,138645  ,274,282.3,289.5
XS GIS Cut Line= 3
2338733.78732315666857.6319508872338957.93991817666825.744479144
2339308.86794322 666630.37022873
#Sta/Elev= 30
       0 2893.06    34.7 2888.22      63 2880.99    71.1 2875.82    79.2 2874.33
   107.5 2861.89   123.6 2856.11   135.7 2853.21   172.1 2838.84   196.3 2827.13
   224.6 2817.09   251.9 2814.12     261 2815.32   283.9 2814.15   297.6 2815.36
   328.5  2815.2   352.6 2811.97     399 2812.69   404.9 2811.55   413.7 2806.53
   421.2 2805.74     435  2805.6   460.8  2805.7   471.6 2806.02   476.2 2807.43
   490.7 2816.87   513.7 2828.88   544.9 2842.18   607.8 2861.17   628.1 2868.55
#Mann= 3 ,-1,0
       0      .1       0   421.2    .045       0   460.8      .1       0
Bank Sta=421.2,460.8
XS Rating Curve= 0 ,0
Exp/Cntr=0.3,0.1

Type RM Length L Ch R = 1 ,138363  ,206.1,214.3,220.1
XS GIS Cut Line= 3
2338818.46131982666961.3817617332338995.50084603 667009.33232213
2339396.11446246666971.891471752
#Sta/Elev= 30
       0 2846.79    22.5 2841.98    88.8 2832.74   126.1 2823.81   170.8 2819.55
   196.1 2815.48   208.2 2815.78   219.4 2813.93   264.4 2812.43   296.6 2812.63
   356.9 2815.44   360.9 2815.17   368.9  2812.6   380.9  2810.7     389 2806.45
     397 2805.28     401 2805.37   436.6 2805.37   441.2 2805.58   445.5  2807.2
   465.3 2824.23   489.4 2838.91   498.6 2846.01   517.5 2858.67   525.6 2862.55
   533.6 2867.54   545.7 2873.45   553.7 2876.25   561.7 2880.65   585.8 2891.64
#Mann= 3 ,-1,0
       0      .1       0     401    .045       0   436.6      .1       0
Bank Sta=401,436.6
XS Rating Curve= 0 ,0
Exp/Cntr(USF)=0,0
Exp/Cntr=0.3,0.1

Type RM Length L Ch R = 1 ,138148  ,222.4,224.1,226.5
XS GIS Cut Line= 3
     2338704.509      667088.6082339085.37522932667161.685170451
2339447.27627966667275.417535586
#Sta/Elev= 30
       0    2831    44.5 2826.79     113 2826.55     130 2822.89   178.9 2817.15
   231.8 2823.16   252.2 2822.85   260.3 2818.49   266.8 2818.25   280.7 2822.79
   309.2 2817.19   325.5 2812.84   338.5 2811.33   427.9 2814.25   436.9 2812.19
   443.9  2809.1   453.6 2807.73   460.1 2805.63   466.2 2804.91   499.8 2805.16
   508.1 2806.49   517.3  2812.4   533.3 2819.59   550.1 2825.77   596.2 2839.25
   646.5 2848.41   667.2 2850.36   709.4 2851.93   756.5 2858.83   767.2 2857.77
#Mann= 5 ,-1,0
       0      .1       0   460.1    .045       0   499.8      .1       0
  537.81     .12       0  637.81      .1       0
Bank Sta=460.1,499.8
XS Rating Curve= 0 ,0
Exp/Cntr=0.3,0.1

Type RM Length L Ch R = 1 ,137924  ,266.6,267.3,268
XS GIS Cut Line= 2
2338598.50005366 667169.913333452339372.11871092667527.553434019
#Sta/Elev= 30
       0 2871.31    76.8 2873.35   116.4 2871.78   136.3 2868.42   147.3 2868.48
   163.4 2863.97   182.5 2860.79   200.1 2855.19   214.7 2846.85   226.6 2842.03
   257.4 2824.49     278  2817.7   288.3 2816.83   332.4 2817.81   345.6 2814.55
   358.8 2816.84   367.6  2814.3   379.5 2812.93   433.7 2813.89   460.1 2810.72
     469 2811.13   477.8 2809.36   486.6 2804.58   494.9 2804.47   537.6 2804.65
   558.2 2812.87   605.6 2815.73   737.8 2834.71   808.5 2842.84   852.3 2846.37
#Mann= 5 ,-1,0
       0      .1       0   486.6    .045       0   537.6      .1       0
     630     .12       0     690      .1       0
Bank Sta=486.6,537.6
XS Rating Curve= 0 ,0
Exp/Cntr(USF)=0,0
Exp/Cntr=0.3,0.1

Type RM Length L Ch R = 1 ,137657  ,224.9,225.8,227.9
XS GIS Cut Line= 3
     2338532.471      667416.751     2338939.009      667621.084
     2339345.548      667825.416
#Sta/Elev= 30
       0 2892.97      40 2892.55    66.8 2889.39    92.5  2881.3   129.5  2855.3
   147.4 2845.46   172.9 2827.44   199.7 2814.84   210.1 2812.77   232.5 2813.19
   245.9  2810.7   299.6 2810.32   317.5 2808.57   326.5 2809.13   344.4 2813.16
   366.6 2811.56   402.6 2811.79   408.3 2811.07   420.2 2804.55     425 2804.25
   475.4 2804.59   492.1 2812.16   496.6 2812.77     590 2815.44   680.1 2816.02
   813.5 2821.33   859.2 2821.83   877.1 2823.65   899.5 2823.09     910 2824.83
#Mann= 4 ,-1,0
       0      .1       0   420.2    .045       0   475.4      .1       0
     775     .12       0
Bank Sta=420.2,475.4
XS Rating Curve= 0 ,0
Exp/Cntr=0.3,0.1

Type RM Length L Ch R = 1 ,137431  ,163.4,166.2,166.1
XS GIS Cut Line= 2
2338448.84923144667626.4751639642339194.56688794667999.333992217
#Sta/Elev= 30
       0 2870.06    13.4 2870.59    41.8 2868.38    52.2 2865.88    58.2 2866.49
    99.9 2856.76     120 2846.73   132.7 2837.37   146.8 2830.97   160.2 2821.38
   173.7 2815.64   186.4 2812.86     205 2810.91   231.8 2810.57   294.4 2812.57
   312.3 2811.37   330.2 2808.07   348.1 2811.67   361.5 2811.69     377 2809.08
     386  2805.4   397.3 2804.12   419.6 2805.67     442  2808.4   450.9 2812.71
   459.9 2813.79     518 2812.23   580.6 2815.49     650 2815.21   833.7 2817.37
#Mann= 5 ,-1,0
       0     .06       0      10      .1       0     386    .045       0
   419.6      .1       0     650     .12       0
Bank Sta=386,419.6
XS Rating Curve= 0 ,0
Exp/Cntr(USF)=0,0
Exp/Cntr=0.3,0.1

Type RM Length L Ch R = 1 ,137265  ,203.8,197.3,193
XS GIS Cut Line= 5
2338443.71253332667863.6047001512338682.82415452667921.638250125
 2338758.4487204667968.1081682032339028.03974806668036.263203284
2339156.37102689 668016.66187638
#Sta/Elev= 30
       0 2845.36    12.8 2846.03    29.3 2845.49    45.8 2843.04    62.2 2837.09
    99.3 2817.34   107.5 2814.53     124  2810.7   144.5 2809.85     161 2810.49
   181.6 2808.12   193.9 2811.08   210.5 2810.47   230.2 2811.33   251.6 2808.79
   261.2 2805.37   266.4 2804.98   298.7 2804.05   306.3 2805.07   319.4 2809.41
   327.5 2813.64   329.2  2813.9   353.1 2812.07   368.8 2813.15   394.4  2811.8
   476.9 2811.42   493.4 2812.04   509.9 2815.18   596.5 2814.64   742.7 2816.47
#Mann= 5 ,-1,0
       0     .06       0     100      .1       0   266.4    .045       0
   306.3      .1       0  612.89     .12       0
Bank Sta=266.4,306.3
XS Rating Curve= 0 ,0
Exp/Cntr=0.3,0.1

Type RM Length L Ch R = 1 ,137068  ,307.5,295.9,288.3
XS GIS Cut Line= 2
2338383.63065242 668057.711432882338947.16256272 668166.63025024
#Sta/Elev= 30
       0    2835    33.1 2832.29    57.6 2831.53    65.7 2830.18      82 2829.43
    95.6 2827.89   105.8 2825.81   118.7 2824.57   126.8  2822.7   147.2 2819.72
   163.5 2814.95     192 2808.65   196.1 2807.46   200.2 2805.39   204.3 2804.79
   233.7 2805.66   257.2 2806.44   269.7 2809.23     302 2812.02   342.8 2812.16
   355.5 2811.54   375.4 2812.67   392.6 2810.14   403.9 2809.52   509.8  2810.2
   513.9 2810.48   525.8  2815.3   530.2 2816.25   554.6 2816.49     574 2815.74
#Mann= 5 ,-1,0
       0      .1       0   200.2    .045       0   233.7      .1       0
     350     .12       0     360      .1       0
Bank Sta=200.2,233.7
XS Rating Curve= 0 ,0
Exp/Cntr(USF)=0,0
Exp/Cntr=0.3,0.1

Type RM Length L Ch R = 1 ,136772  ,271.1,259.9,252.9
XS GIS Cut Line= 3
2338349.70139518668406.8362167652338590.74411644 668416.62916029
2338988.16693529668230.155806292
#Sta/Elev= 30
       0 2841.62    66.9 2837.37   130.6  2830.4   154.6 2828.72   166.6 2826.47
   178.6 2826.65   190.6 2824.09   218.7 2821.56   241.2 2815.42   269.3 2809.41
     287 2811.06     293 2808.93   300.3  2804.5     312 2803.56   313.5 2803.54
   338.1 2803.64   359.2 2804.63   368.2 2809.13   380.2 2810.86   401.3 2810.35
   410.7 2811.56   425.4 2811.61   516.8 2810.23     530 2809.28   552.1 2809.99
   617.8 2809.31   632.9 2809.96   644.9 2814.38   650.9  2815.7   680.2 2815.82
#Mann= 5 ,-1,0
       0     .06       0     190     .12       0     312    .045       0
   338.1     .12       0  401.24      .1       0
Bank Sta=312,338.1
XS Rating Curve= 0 ,0
Exp/Cntr=0.3,0.1

Type RM Length L Ch R = 1 ,136512  ,152.3,150,150.2
XS GIS Cut Line= 2
2338775.10370062668709.4217685332338999.60638618668234.653794159
#Sta/Elev= 30
       0  2836.4     4.7 2837.29    57.8 2840.54    88.8 2840.29   106.5 2839.03
   121.2 2834.97   127.2 2832.23   150.7 2815.15   155.1 2812.83   170.9 2809.63
   184.2 2809.05   199.4 2804.21   205.3  2803.1   208.2 2803.06   241.7 2803.12
   252.5 2804.47   261.3 2806.97   270.2 2807.05   292.3    2810     310  2809.3
     330 2810.97   354.2 2810.09   398.5 2810.17   438.3 2808.75   466.6  2809.1
   478.1 2810.08     487 2814.18   491.4 2815.09   504.7 2815.94   525.2 2815.32
#Mann= 5 ,-1,0
       0     .06       0     130      .1       0   205.3    .045       0
   241.7     .12       0     330      .1       0
Bank Sta=205.3,241.7
XS Rating Curve= 0 ,0
Exp/Cntr(USF)=0,0
Exp/Cntr=0.3,0.1

Type RM Length L Ch R = 1 ,136362  ,260.4,258.2,253.2
XS GIS Cut Line= 2
2338852.87344018669000.867200076 2339162.5366235668134.506159092
#Sta/Elev= 30
       0 2825.56    20.9 2825.71    45.5 2828.38    71.2 2828.95   101.6 2825.32
   110.1 2828.79   148.3 2832.57   284.3  2835.4   335.2 2839.63   360.7 2840.25
   373.5 2836.13   394.7 2820.76   411.7 2811.53   421.7 2809.14   437.2 2808.97
   445.7 2806.57   458.4 2806.42     470 2803.57   481.1 2802.94   515.5 2803.62
   534.9 2809.34   564.6 2808.64     575 2810.27   590.1 2810.41   628.3 2808.34
   703.3 2808.67     719 2814.53   734.5 2815.37   819.5 2813.62     920  2814.6
#Mann= 7 ,-1,0
       0     .12       0     210      .1       0     310     .06       0
     410      .1       0     470    .045       0   515.5      .1       0
     830     .12       0
Bank Sta=470,515.5
XS Rating Curve= 0 ,0
Exp/Cntr(USF)=0,0
Exp/Cntr=0.3,0.1

Type RM Length L Ch R = 1 ,136104  ,211.8,211.9,212.7
XS GIS Cut Line= 3
 2339081.4251666669550.5638775362339280.50906144668503.662877111
 2339355.0974932668149.806565809
#Sta/Elev= 30
       0 2835.48    89.1 2833.31   103.2 2834.03   119.5  2830.7   229.4 2818.27
   274.2 2815.39   347.5 2814.42   355.6 2811.18   367.9 2809.89   407.2 2809.37
   445.2 2811.65   482.5 2808.84   754.7 2808.76   811.7 2809.44   823.9 2811.44
     885 2804.97   929.8 2802.88   974.5 2802.76   975.1 2802.93   982.7 2806.19
   994.9  2805.3  1015.3 2807.22  1035.6 2806.14  1051.9 2809.26  1083.4 2807.93
  1121.3 2808.24  1162.2 2813.79  1198.8 2813.98  1227.6 2812.27  1427.3 2818.66
#Mann= 10 ,-1,0
       0     .06       0      60      .1       0     460     .12       0
     560      .1       0     750    .025       0     860      .1       0
   929.8    .045       0   975.1      .1       0 1155.66     .06       0
 1255.66      .1       0
#XS Ineff= 2 , 0
          823.06 2816.78
Permanent Ineff=
       T       F
Bank Sta=929.8,975.1
XS Rating Curve= 0 ,0
Exp/Cntr=0.3,0.1

Type RM Length L Ch R = 1 ,135892  ,332,340.1,353.9
XS GIS Cut Line= 3
2339350.42215046669195.7114502572339500.03469971668468.524873688
2339580.06001675668172.779136806
#Sta/Elev= 30
       0 2825.41    27.1 2821.99    43.4 2818.33   108.8 2815.09   125.6  2812.7
   152.7  2812.6   161.9 2809.53     438 2808.75     460  2811.2   476.3 2806.13
   488.6 2804.21   521.8 2804.46   544.6 2807.95     558 2805.35   570.2 2805.08
   576.9 2803.08   582.5 2802.66   623.1  2803.2   631.5 2805.97   639.7 2806.48
   651.9 2805.73   660.1 2806.92   703.4 2806.11     750 2807.27   762.5 2809.04
   774.6 2812.83   791.5 2814.24   890.9 2814.34   977.9 2819.78  1048.8 2821.83
#Mann= 8 ,-1,0
       0     .06       0     100      .1       0     200    .025       0
     500      .1       0   576.9    .045       0   623.1      .1       0
  802.42     .06       0 1002.42      .1       0
#XS Ineff= 2 , 0
          457.89 2814.13
Permanent Ineff=
       T       F
Bank Sta=576.9,623.1
XS Rating Curve= 0 ,0
Exp/Cntr(USF)=0,0
Exp/Cntr=0.3,0.1

Type RM Length L Ch R = 1 ,135552  ,246.6,246.5,246.4
XS GIS Cut Line= 5
2339527.53730154 669098.628238692339562.84455064668819.002192958
2339703.64733593 668708.262106222339914.01570392668552.485053686
2339965.51673151668531.674517678
#Sta/Elev= 30
       0 2815.03    94.2 2815.04   106.3  2815.9   122.4 2812.51   213.1 2810.76
   283.5 2811.81   324.3 2810.86   346.8 2809.26   362.4 2809.49   369.5 2808.31
   407.7 2806.01   466.2 2805.78   480.7 2806.31   503.6 2808.84   519.9 2805.67
   536.3 2804.23   551.2 2804.24   560.3 2802.28   566.2  2802.1   580.4 2802.04
   600.8 2802.06   606.5 2802.27   623.7 2805.39   660.7 2806.56   669.5 2810.23
   685.6    2813   706.6 2824.04   723.9 2828.47   742.3 2824.24   778.3 2822.64
#Mann= 6 ,-1,0
       0      .1       0     100    .025       0     190      .1       0
   566.2    .045       0   600.8      .1       0  720.98     .06       0
#XS Ineff= 2 , 0
          502.88 2813.98
Permanent Ineff=
       T       F
Bank Sta=566.2,600.8
XS Rating Curve= 0 ,0
Exp/Cntr=0.3,0.1

Type RM Length L Ch R = 1 ,135305  ,186.5,191.6,202.4
XS GIS Cut Line= 3
2339578.46210397669134.9157866732340062.12496543668737.744732125
2340526.30510647668603.866914356
#Sta/Elev= 30
       0 2816.79    48.8 2816.17   126.4 2817.86   152.3 2809.88   311.6  2809.9
   329.3 2811.92   349.4 2809.52     437 2807.71   494.4 2801.96   513.3 2801.41
   542.4 2801.96     551 2804.92   592.3 2839.24   614.1 2852.32   702.9 2887.13
     732 2895.51   765.4 2897.17     807 2894.15   815.4 2891.48   827.8 2883.61
   858.8 2873.91   873.5 2870.19   881.9 2869.49   898.6 2864.13   915.2 2861.54
   931.9  2856.8   951.1 2855.86   990.2 2851.34    1011 2852.73  1108.9  2850.5
#Mann= 5 ,-1,0
       0     .07       0      50      .1       0   494.4    .045       0
   542.4     .06       0  675.84      .1       0
#XS Ineff= 2 , 0
             329 2817.71
Permanent Ineff=
       T       F
Bank Sta=494.4,542.4
XS Rating Curve= 0 ,0
Exp/Cntr(USF)=0,0
Exp/Cntr=0.3,0.1

Type RM Length L Ch R = 1 ,135114  ,280.6,288.4,293.7
XS GIS Cut Line= 3
 2339561.7737018669201.7021272472339793.26166585669081.331741624
2340224.53336765668921.845188928
#Sta/Elev= 30
       0 2819.91    52.3 2817.89   147.5 2820.23   180.1 2820.11   192.1 2819.32
   196.6 2818.24   212.8 2811.31   218.7 2809.89     345 2809.88   353.6 2811.35
   362.1 2811.63   374.9  2809.5   387.7 2808.53   428.3  2807.5   464.5 2808.03
   481.5 2806.51   490.6 2802.64   498.6 2801.34     537 2800.94   543.5 2801.03
   559.1  2804.4   583.6 2824.76   609.5 2839.52     618 2845.33   626.5  2852.4
   639.3 2860.09   652.5 2865.46   669.2 2874.77   688.1 2882.63   720.7 2899.68
#Mann= 8 ,-1,0
       0     .07       0      70      .1       0  280.91    .025       0
  470.91      .1       0   498.6    .045       0   543.5      .1       0
  600.91     .06       0  700.91      .1       0
Bank Sta=498.6,543.5
XS Rating Curve= 0 ,0
Exp/Cntr=0.3,0.1

Type RM Length L Ch R = 1 ,134825  ,182.1,184.6,189.1
XS GIS Cut Line= 2
2339542.96508981669298.1354123282340220.95940813669261.610465887
#Sta/Elev= 30
       0 2834.59    13.2 2831.36    29.3 2828.79    57.3 2821.87    81.3 2818.93
   105.4 2818.48   121.4 2819.57   181.5 2820.38   197.5 2821.48   237.6 2820.59
   249.6 2817.94   261.6 2816.68   273.6 2809.89   381.8 2809.88   397.8 2810.56
   405.8 2808.92   417.8 2808.21   425.8 2805.72   454.4 2800.33   461.8 2799.97
   501.9 2800.03   507.6 2801.59     514 2804.56     522  2810.4     530 2815.16
     570 2844.25   590.1 2855.63   638.1 2886.04     652 2894.06     679 2907.79
#Mann= 5 ,-1,0
       0      .1       0     370    .025       0   454.4    .045       0
   501.9     .06       0     670      .1       0
Bank Sta=454.4,501.9
XS Rating Curve= 0 ,0
Exp/Cntr(USF)=0,0
Exp/Cntr=0.3,0.1

Type RM Length L Ch R = 1 ,134641  ,258.6,257.7,257.1
XS GIS Cut Line= 2
     2339541.288      669425.4422340183.13983681669466.608447304
#Sta/Elev= 30
       0 2835.62    18.9 2829.19      31 2827.09    95.1 2822.14   127.1 2818.07
   151.2 2817.66   167.2 2815.73   223.3 2812.08   263.4 2810.43   287.5 2811.42
   307.5 2807.21   322.6 2805.99   355.6 2806.08   386.7 2807.54   399.7 2805.34
     413 2800.39   424.3 2799.41   459.8 2799.29   461.6  2799.3   475.9 2799.57
   483.9  2802.7   495.9  2805.5   508.8 2811.41     524 2819.75     540 2831.76
     552 2838.84   576.1 2857.73   600.1 2874.18   620.8 2885.69   643.2 2894.63
#Mann= 5 ,-1,0
       0      .1       0   424.3    .045       0   461.6      .1       0
     470     .06       0     570      .1       0
#XS Ineff= 2 , 0
          383.04 2822.66
Permanent Ineff=
       F       F
Bank Sta=424.3,461.6
XS Rating Curve= 0 ,0
Exp/Cntr=0.3,0.1

Type RM Length L Ch R = 1 ,134383  ,222,225.3,226.6
XS GIS Cut Line= 2
2339356.41997618669677.1943169232340155.38449411669720.149398532
#Sta/Elev= 30
       0 2845.65    51.8 2843.83    71.9 2841.95   131.9 2831.48     152 2823.79
     156 2822.83     164 2822.82     176 2818.62   212.1 2810.98   316.2 2810.56
   356.3 2811.99   389.2  2811.1   420.4 2812.13   428.4 2810.98   480.4 2808.18
   508.5 2804.77   536.5 2806.55   552.6 2802.84   560.6 2799.27     570 2798.69
   584.6  2798.6   623.2 2798.79   628.7 2799.55   648.7    2806   680.7 2826.19
   704.8 2837.86   728.8 2845.69     760  2853.4   768.9 2854.84   800.1 2862.98
#Mann= 9 ,-1,0
       0      .1       0      70     .06       0     390     .12       0
     460     .06       0     560      .1       0     570    .045       0
   623.2      .1       0     660     .06       0     760      .1       0
Bank Sta=570,623.2
XS Rating Curve= 0 ,0
Exp/Cntr(USF)=0,0
Exp/Cntr=0.3,0.1

Type RM Length L Ch R = 1 ,134158  ,233.7,234.1,232.9
XS GIS Cut Line= 3
2339205.71302852669851.0032559312339511.33560676669873.177853104
2340150.70251666669963.950597172
#Sta/Elev= 30
       0 2833.58    10.5  2833.3    30.5 2834.25    70.6 2830.96   191.3 2826.86
     215 2823.66   243.1 2816.62   254.9 2815.34   279.2 2810.04   400.2 2809.38
   472.9 2810.35   545.6 2809.29   553.7 2808.79   569.9 2805.45     578 2804.68
   598.2 2804.45   607.9 2805.63   653.9 2805.38     679 2801.71   691.1 2798.65
   698.2 2798.09   706.9    2798   747.6 2798.28     784 2806.39   796.1  2808.5
   804.2 2808.73   827.2 2812.96   912.1 2822.54   921.4 2822.48   952.2 2824.74
#Mann= 8 ,-1,0
       0      .1       0      20     .06       0     120      .1       0
     220     .12       0  516.43     .06       0   698.2    .045       0
   747.6     .06       0  816.43      .1       0
Bank Sta=698.2,747.6
XS Rating Curve= 0 ,0
Exp/Cntr=0.3,0.1

Type RM Length L Ch R = 1 ,133924  ,142.2,140.9,140.2
XS GIS Cut Line= 3
2339197.48617422670080.9720840532340000.74620032670175.473263594
2340176.86203492670089.563100375
#Sta/Elev= 30
       0 2819.38    14.8 2816.87    34.9 2815.66   111.5 2812.84   147.7 2813.75
   216.2 2811.14   256.4 2811.58   280.1 2810.36   300.7 2807.09   369.2  2804.8
     486 2803.51   507.1 2800.62   518.2 2801.59   530.3 2800.22   538.4 2803.32
     631 2803.93   659.2 2798.22   675.3 2797.16   679.3 2797.13   715.6 2797.21
   723.6 2800.28   730.5 2801.39   747.8 2801.34   763.9 2803.43     780 2802.57
   808.8 2806.53     826 2807.27   935.7 2809.35   965.6 2814.21  1004.8 2817.27
#Mann= 8 ,-1,0
       0      .1       0     100     .12       0     430     .06       0
     620     .12       0   675.3    .045       0   715.6     .12       0
   818.8     .06       0   928.8     .12       0
#XS Ineff= 2 , 0
          457.13 2809.05
Permanent Ineff=
       F       F
Bank Sta=675.3,715.6
XS Rating Curve= 0 ,0
Exp/Cntr(USF)=0,0
Exp/Cntr=0.3,0.1

Type RM Length L Ch R = 1 ,133783  ,152.6,148,143.9
XS GIS Cut Line= 3
 2339363.3555269670266.3301391782340063.19203983670315.038647402
 2340205.4475043670245.493824331
#Sta/Elev= 30
       0 2812.32     8.8 2809.65    16.9 2809.21   108.4 2807.99   117.1    2807
   125.1 2807.82   142.1 2811.98   157.2 2812.94   197.3 2811.01   217.3 2803.82
   265.5 2803.85   273.6 2802.37   285.5 2802.07   393.8 2800.87   421.8 2803.55
     446  2804.4   468.3  2801.4     478  2796.6     482 2796.57   530.1 2796.41
   549.4 2796.62   558.2 2799.55   586.2 2804.12   602.3  2803.8   618.3 2805.95
   646.4 2807.02     805 2807.39   820.3 2809.26   831.7 2809.17   859.9  2812.6
#Mann= 6 ,-1,0
       0      .1       0      60     .12       0     360     .06       0
     482    .045       0   549.4     .06       0     650     .12       0
#XS Ineff= 2 , 0
                          715.59         2808.63
Permanent Ineff=
       F       F
Bank Sta=482,549.4
XS Rating Curve= 0 ,0
Exp/Cntr=0.3,0.1

Type RM Length L Ch R = 1 ,133635  ,508,505.3,476.3
XS GIS Cut Line= 3
2339298.60799152670487.1732925042340068.73633353670438.381479676
 2340272.2217417670248.927823417
#Sta/Elev= 30
       0 2819.18    25.6 2819.46   113.8 2816.11   173.9 2815.16     194 2810.63
   203.1  2806.3     218 2803.16   270.1  2802.8   302.2 2804.31   358.3 2803.77
   374.3  2801.9   398.4 2801.94   418.4 2803.12   470.5 2800.15   518.6 2802.51
   549.9 2796.12   550.7 2796.03     614 2796.31   618.8 2797.67   630.8 2803.94
   646.9 2805.59   666.7 2805.23   686.9  2806.7   777.8 2805.91   947.6 2807.75
   961.8 2808.52   990.6 2812.94  1014.1 2813.73  1025.9 2815.34  1049.7 2815.62
#Mann= 5 ,-1,0
       0     .12       0     420     .06       0   549.9    .045       0
     614     .06       0  831.67     .12       0
#XS Ineff= 2 , 0
                          842.84          2808.3
Permanent Ineff=
       F       F
Bank Sta=549.9,614
XS Rating Curve= 0 ,0
Exp/Cntr(USF)=0,0
Exp/Cntr=0.3,0.1

Type RM Length L Ch R = 1 ,133130  ,325.9,312.5,282.6
XS GIS Cut Line= 3
 2339448.0579401671096.9760895592339774.68214946670890.807245864
2340360.39442746670313.577099322
#Sta/Elev= 30
       0 2845.43    52.2 2843.46    85.3 2836.77   104.5 2830.56   127.9 2825.15
   146.8 2827.19   170.4 2826.15   198.8 2818.45   227.2 2807.07   231.9 2807.72
   246.9 2816.52   255.6 2817.72   276.9 2805.42   310.2 2798.84   318.9 2796.65
   378.6 2799.19   405.4 2802.18   444.5 2801.86   464.8  2803.5   489.4 2803.63
   518.6 2801.02   570.9  2804.3     588 2803.72   629.8 2805.89   713.7 2805.77
   767.5 2803.15   809.5 2806.34   835.4 2804.86   998.3 2806.28  1208.6 2811.45
#Mann= 7 ,-1,0
       0      .1       0   310.2    .045       0   378.6      .1       0
  446.25     .12       0  586.25      .1       0  826.25     .06       0
  966.25     .12       0
#XS Ineff= 2 , 0
                          964.26         2808.66
Permanent Ineff=
       F       F
Bank Sta=310.2,378.6
XS Rating Curve= 0 ,0
Exp/Cntr=0.3,0.1

Type RM Length L Ch R = 1 ,132817  ,188.7,187.1,185.7
XS GIS Cut Line= 4
 2339853.9158305671466.647237984   2340084.16396 670852.22110786
2340170.54689428670538.5397302532340386.57129943670329.556583771
#Sta/Elev= 30
       0 2845.03    22.9 2846.13   108.5 2856.21   155.3 2859.82   159.6 2859.16
     181 2862.31     208 2864.11   236.5 2864.13   282.5  2861.3   350.9 2851.31
   368.9 2846.19   381.7 2840.58   390.3 2838.99   407.4 2829.69     433 2820.24
   453.4 2803.55   465.9 2797.53   472.1 2795.76   488.5 2795.57   514.2 2795.66
   534.2 2797.96   544.1 2801.27   569.7 2803.31   642.3 2804.98   680.1 2802.55
   707.4 2803.94   870.9 2803.77   895.8 2805.24  1082.6 2806.38  1282.1  2811.7
#Mann= 7 ,-1,0
       0      .1       0   465.9    .045       0   534.2      .1       0
     630     .12       0  736.15      .1       0  936.15     .06       0
 1061.51     .12       0
Bank Sta=465.9,534.2
XS Rating Curve= 0 ,0
Exp/Cntr(USF)=0,0
Exp/Cntr=0.3,0.1

Type RM Length L Ch R = 1 ,132630  ,242.7,234.3,229
XS GIS Cut Line= 3
2339983.76629598671727.2440304592340158.03896349 671219.84678722
2340421.27696349670331.927265831
#Sta/Elev= 30
       0 2853.53   120.6 2855.05   188.3 2851.96   260.2 2851.16   277.1  2849.5
   315.2 2852.02     404  2850.3   445.8 2854.32   475.9 2854.74   508.8 2852.58
   546.8 2845.43   572.9 2837.99   611.2  2823.1   635.2  2808.1   656.2 2802.22
   669.1 2801.78   681.1 2796.94     702 2795.69   722.8 2796.75   739.5 2796.79
   777.1  2803.1   818.8 2800.01   856.4 2803.29   923.1 2801.98   989.9  2804.3
  1023.2 2802.99  1203.3 2804.38  1306.2 2807.67  1394.6 2808.41  1462.6 2812.43
#Mann= 8 ,-1,0
       0      .1       0   681.1    .045       0   722.8      .1       0
  796.49     .12       0  896.49      .1       0 1056.49     .08       0
 1106.49     .06       0 1306.49     .12       0
Bank Sta=681.1,722.8
XS Rating Curve= 0 ,0
Exp/Cntr=0.3,0.1

Type RM Length L Ch R = 1 ,132396  ,256.5,248.2,239.2
XS GIS Cut Line= 3
 2340466.3018587671684.4677317672340423.34677709670705.091871069
2340436.13162354670358.116040858
#Sta/Elev= 30
       0 2815.35    47.3 2813.25   112.6 2812.33   167.4 2807.44   207.5 2807.76
   235.7 2809.74   252.5 2812.73   323.5 2809.84   347.6 2811.03   383.7 2810.59
   423.7 2814.22   535.8 2818.03   551.8 2817.23   559.8 2815.54   567.8 2811.75
   575.8 2805.86   611.9 2796.21   639.9 2795.45   649.6 2796.08   655.9 2799.53
   671.9 2801.99     700 2800.04     712 2802.39     736 2803.15     792 2801.34
  1032.3 2802.46  1136.3 2804.75  1180.4 2807.33  1232.4  2806.8  1327.5 2809.16
#Mann= 9 ,-1,0
       0      .1       0     520     .12       0   611.9    .045       0
   649.6     .12       0     710      .1       0     810     .12       0
     910     .08       0 1010.32     .06       0 1110.32     .12       0
Bank Sta=611.9,649.6
XS Rating Curve= 0 ,0
Exp/Cntr(USF)=0,0
Exp/Cntr=0.3,0.1

Type RM Length L Ch R = 1 ,132147  ,238,244,253.9
XS GIS Cut Line= 4
2340727.31701581671138.6485964022340660.07374687670958.527733291
2340605.86947009 670857.87484813 2340607.1821267670399.024788692
#Sta/Elev= 30
       0 2840.51    14.4 2837.76    27.2 2836.71    61.3 2830.64    81.3 2828.63
   108.3  2824.4   138.2 2816.92   155.3 2815.35   180.9 2810.36   193.8 2806.65
     202 2802.42   222.7 2794.84   243.8 2794.15   257.4 2795.04     271 2798.19
   307.3 2801.79   351.3 2799.89   443.3 2799.26   463.3 2799.94   543.3 2799.97
   555.3 2801.01   579.3 2800.19   611.3 2801.02   639.3  2803.7   655.3 2808.97
   659.3 2809.63   691.3 2811.82   735.3 2812.31   743.3 2813.33   765.4 2813.99
#Mann= 8 ,-1,0
       0      .1       0     180     .12       0   222.7    .045       0
   257.4     .12       0  292.26      .1       0  486.58     .12       0
  586.58     .06       0  686.58      .1       0
Bank Sta=222.7,257.4
XS Rating Curve= 0 ,0
Exp/Cntr=0.3,0.1

Type RM Length L Ch R = 1 ,131903  ,314.5,331.2,346.1
XS GIS Cut Line= 4
2340776.17874355671153.9985046682340867.49110965670869.915587905
2340766.03292509670608.660762666 2340804.0797443670362.624665112
#Sta/Elev= 30
       0 2842.61     9.3 2839.43    51.3 2832.74    70.6 2826.46      96 2823.35
   122.7 2815.17   164.7 2806.92   210.9  2800.8   240.3 2800.28   265.6 2803.03
   346.4 2803.09     355 2801.56   375.7 2794.08   384.9 2793.62   440.6 2793.53
   455.2 2793.59   462.3 2793.88   470.8  2797.9   483.9 2801.42   530.9 2799.18
   558.1 2796.32   582.2 2798.99   614.6 2799.94   630.8 2802.78   646.9 2807.48
     676 2809.97   695.5 2809.28   715.8 2811.78     740 2818.91   827.6 2835.43
#Mann= 6 ,-1,0
       0      .1       0     290     .12       0   384.9    .045       0
   455.2     .12       0  608.66     .06       0  708.66      .1       0
Bank Sta=384.9,455.2
XS Rating Curve= 0 ,0
Exp/Cntr(USF)=0,0
Exp/Cntr=0.3,0.1

Type RM Length L Ch R = 1 ,131572  ,240.5,252.2,266.3
XS GIS Cut Line= 4
2340820.42726309671199.0011814822341056.59356797670921.602145489
2341080.35050792670752.0522448272341177.61219489  670383.3579659
#Sta/Elev= 30
       0 2844.29    39.2 2836.29    55.1  2830.2    66.4 2828.39    91.9 2819.33
   108.9 2815.46   179.9 2804.68   364.3 2803.56   409.2 2799.26   433.4 2798.45
   485.9 2801.82   581.9 2802.27   608.8 2800.67   629.5 2797.37   637.8 2794.76
   678.5 2793.29   691.6 2794.75   691.6 2794.76   691.6  2794.8     704 2802.16
   724.6 2807.43   741.2 2819.89   757.7  2827.9     795 2838.76   807.4 2844.92
   819.8  2848.8   832.2 2855.68   840.5 2857.94   881.8 2876.38   916.8 2890.28
#Mann= 5 ,-1,0
       0      .1       0  615.52     .06       0   637.8    .045       0
   691.6     .06       0  715.52      .1       0
#XS Ineff= 2 , 0
          213.68 2822.51
Permanent Ineff=
       F       F
Bank Sta=637.8,691.6
XS Rating Curve= 0 ,0
Exp/Cntr=0.3,0.1

Type RM Length L Ch R = 1 ,131320  ,179.1,179,184
XS GIS Cut Line= 2
2340867.88468511671233.4295854032341434.02135495670651.313251499
#Sta/Elev= 30
       0  2839.6    17.1 2836.64    29.1 2832.66    42.8 2825.99    61.7 2821.58
     122 2812.67   134.3 2811.71   172.5 2804.07   418.8 2801.96   459.4  2797.3
   488.1 2799.98   532.2 2800.29   546.3 2798.66   560.5 2799.81   591.4 2796.95
   600.1 2794.38   608.5 2793.34     617 2793.24   631.5 2793.29     643  2794.1
   647.6 2795.68   658.8 2806.35   677.4  2812.6   688.9 2820.52   704.7 2833.77
     750 2851.65   757.7 2856.15   770.4 2859.42   781.5 2864.97     812 2874.28
#Mann= 4 ,-1,0
       0      .1       0   608.5    .045       0   631.5      .1       0
     750     .06       0
#XS Ineff= 2 , 0
          212.55  2819.7
Permanent Ineff=
       F       F
Bank Sta=608.5,631.5
XS Rating Curve= 0 ,0
Exp/Cntr(USF)=0,0
Exp/Cntr=0.3,0.1

Type RM Length L Ch R = 1 ,131141  ,250,246.7,249.3
XS GIS Cut Line= 3
 2340851.0180341671297.5149025552341258.90911571671017.443228991
2341584.28852618670837.387081609
#Sta/Elev= 30
       0 2856.41    71.3 2834.27    87.4 2826.32   214.9 2806.09   234.3 2804.33
   258.6 2803.81   326.5 2803.91   354.9 2802.76   455.6  2802.2   534.2 2797.84
   555.7 2799.51     574 2799.64     593  2798.1   596.8 2797.06   601.4 2793.93
   604.8  2793.1   640.1 2792.92   642.5 2792.92   656.2 2796.66   675.4 2807.61
   690.2 2810.26   697.4 2814.83   706.5 2823.56   711.1 2826.91   724.8 2831.45
   738.5 2834.57   752.2 2839.19   796.1  2851.2   825.4 2857.27   866.7 2871.28
#Mann= 5 ,-1,0
       0      .1       0   604.8    .045       0   642.5      .1       0
  754.79     .06       0  866.66      .1       0
#XS Ineff= 2 , 0
           386.8 2806.26
Permanent Ineff=
       F       F
Bank Sta=604.8,642.5
XS Rating Curve= 0 ,0
Exp/Cntr=0.3,0.1

Type RM Length L Ch R = 1 ,130894  ,171,179.5,181
XS GIS Cut Line= 2
2341050.28882579671419.6171838982341726.00033495671026.974009656
#Sta/Elev= 30
       0 2839.19    20.7 2830.08    28.7 2828.56    35.3 2825.37    70.5 2814.98
      88 2813.35   102.6 2809.95   117.3 2809.54     141 2806.15   187.5 2802.16
   293.6 2802.77   353.8 2798.73   383.5 2798.46   427.4 2792.34   450.7 2792.16
   464.8 2792.34   483.3 2796.07   498.5 2804.14   518.1  2804.3   529.8 2810.27
   550.6 2814.78   575.8 2819.23   608.9 2822.35   641.8 2827.98   659.1  2833.1
   711.3 2845.27     723 2849.21   729.4 2849.19   766.9 2857.22   781.5 2861.44
#Mann= 5 ,-1,0
       0      .1       0   427.4    .045       0   464.8      .1       0
     620     .06       0     740      .1       0
#XS Ineff= 2 , 0
          241.49 2816.13
Permanent Ineff=
       F       F
Bank Sta=427.4,464.8
XS Rating Curve= 0 ,0
Exp/Cntr(USF)=0,0
Exp/Cntr=0.3,0.1

Type RM Length L Ch R = 1 ,130715  ,244.2,229.1,221.3
XS GIS Cut Line= 4
2341220.43973323671487.3835150312341312.06104239671412.590609593
2341611.23266414671328.4485909742341753.33918448671193.821361185
#Sta/Elev= 30
       0 2826.31    30.6  2811.8      41  2808.5    46.9 2807.64    61.6 2807.68
   117.3 2802.96   143.3 2803.64   155.8 2802.42   180.7 2797.15   222.3 2799.02
   231.4 2798.11     243 2795.49   259.7 2795.04   281.2 2791.73   299.5 2791.62
   328.7 2791.69   338.6  2792.5   346.9 2797.06   367.3 2796.46   380.2 2800.36
   405.1 2800.55   421.7 2803.11   468.7 2806.38   485.4 2808.53   507.5 2806.83
   555.9 2814.49   568.1 2815.04   579.1 2817.61   606.7 2820.66   624.8  2825.1
#Mann= 3 ,-1,0
       0      .1       0   281.2    .045       0   328.7      .1       0
Bank Sta=281.2,328.7
XS Rating Curve= 0 ,0
Exp/Cntr(USF)=0,0
Exp/Cntr=0.3,0.1

Type RM Length L Ch R = 1 ,130486  ,158.1,149.1,147
XS GIS Cut Line= 3
2341407.60716038671753.8626460042341720.45788489671413.508858486
2341817.02721608671263.410813155
#Sta/Elev= 30
       0 2877.16    22.7 2873.26    33.5 2870.07    42.2 2869.33    77.7 2855.56
    85.8 2853.45    95.4 2852.35   128.3 2840.14   142.2 2833.92   153.8 2830.51
   169.4 2822.63   184.1 2811.73   201.8 2800.51   219.5 2792.06   231.4 2791.44
   260.9 2791.57   267.2 2791.87   281.1  2794.9     301 2796.57   314.1 2796.44
   332.1 2797.77   343.7 2799.73   379.1 2800.15   408.4 2801.57   426.4  2801.1
   502.8 2803.41     534 2805.23   540.5 2806.08   557.8 2810.75   640.8 2827.07
#Mann= 4 ,-1,0
       0      .1       0   219.5    .045       0   260.9      .1       0
  582.29     .06       0
Bank Sta=219.5,260.9
XS Rating Curve= 0 ,0
Exp/Cntr=0.3,0.1

Type RM Length L Ch R = 1 ,130337  ,185,179.2,169.8
XS GIS Cut Line= 2
2341607.72948676671846.1202428642341876.59367584671288.100227792
#Sta/Elev= 30
       0  2841.9    23.2 2839.22    36.6 2839.75    58.8 2838.02    75.9 2838.47
    98.7 2837.41   129.9 2834.33     152 2829.53   165.8 2824.49   194.5 2800.52
   198.8  2797.7   210.8 2793.11   216.8 2791.73   249.7 2791.34   264.7 2791.59
   305.1 2799.47   360.6 2800.12   396.6 2801.54   406.5 2800.89   431.7 2802.01
   480.6 2802.15   513.4 2807.81     525 2808.46   535.5 2811.16   546.4 2812.19
   556.1 2814.35   564.9 2814.76   582.7 2820.13   591.6 2820.77   619.4 2828.24
#Mann= 4 ,-1,0
       0      .1       0   216.8    .045       0   264.7      .1       0
     530     .06       0
Bank Sta=216.8,264.7
XS Rating Curve= 0 ,0
Exp/Cntr(USF)=0,0
Exp/Cntr=0.3,0.1

Type RM Length L Ch R = 1 ,130157  ,249.9,255.7,259.7
XS GIS Cut Line= 3
2341851.36553084671942.597727535 2341899.6821491 671559.45966197
2341971.74176736671270.310785334
#Sta/Elev= 30
       0 2851.45    65.3 2841.17   110.3 2830.27   126.4    2829   199.1 2818.22
   231.4 2808.69   239.3 2803.58   259.5  2792.8   272.9 2791.23   287.7 2790.96
   320.6  2791.2     328 2791.58   336.1 2795.05   344.1 2795.81   356.2 2799.21
   377.9 2801.27   400.9 2800.53   431.4 2801.72   466.8 2799.98   499.8 2801.52
   524.6 2805.05     541 2805.33     574 2813.44   590.5  2819.7   598.8 2819.24
     607 2824.06   615.3 2827.17   668.8  2844.2   677.1 2845.16   684.2 2847.31
#Mann= 4 ,-1,0
       0      .1       0   272.9    .045       0   320.6      .1       0
  586.17     .06       0
#XS Ineff= 2 , 0
                          431.71         2810.31
Permanent Ineff=
       F       F
Bank Sta=272.9,320.6
XS Rating Curve= 0 ,0
Exp/Cntr=0.3,0.1

Type RM Length L Ch R = 1 ,129902  ,272.4,285.2,293.7
XS GIS Cut Line= 3
2341929.85922273671995.7710650882342120.09331878671724.370421394
2342236.77023102 671427.60523156
#Sta/Elev= 30
       0 2851.47    22.7 2846.75    37.4 2842.49      52 2840.08    61.8 2836.49
   101.6 2829.47   149.7 2822.57   164.3 2818.72     179  2816.9   208.3 2810.95
   221.8 2809.55   252.3 2803.89   289.8 2801.16   320.7  2796.9   339.2 2795.98
     371 2790.14   407.9 2789.84   412.2 2790.04   429.4 2791.69   441.9 2799.45
   446.6 2801.25   460.4 2799.83   472.4 2803.95   489.6 2805.06     516 2809.82
   554.1 2822.44   584.1 2836.32   596.2 2839.76   618.5 2851.57   650.3 2864.65
#Mann= 4 ,-1,0
       0      .1       0     371    .045       0   412.2     .06       0
  501.43      .1       0
#XS Ineff= 2 , 0
                          446.75         2809.96
Permanent Ineff=
       F       F
Bank Sta=371,412.2
XS Rating Curve= 0 ,0
Exp/Cntr(USF)=0,0
Exp/Cntr=0.3,0.1

Type RM Length L Ch R = 1 ,129617  ,319.3,319.2,299.1
XS GIS Cut Line= 2
2342000.64101027672124.8774249822342443.83678095671777.313993152
#Sta/Elev= 30
       0 2880.44    25.4 2872.17    44.9 2868.48    57.8 2861.53    70.7 2860.03
    77.3 2857.79   136.7 2834.64     159 2822.46     168 2821.26   182.4 2813.48
   192.6 2810.66   201.7  2806.1     218 2801.89   243.4 2800.51   268.8 2801.35
   290.1 2799.36   315.7 2799.16   358.4 2795.19   381.9 2795.76     401 2790.49
   407.9 2790.08   431.5 2789.51   433.8 2789.51   453.3 2790.58   467.1 2797.84
   482.3 2802.15   486.6 2805.35   507.7 2826.07   517.9 2832.68   563.2 2845.18
#Mann= 3 ,-1,0
       0      .1       0   407.9    .045       0   433.8     .06       0
Bank Sta=407.9,433.8
XS Rating Curve= 0 ,0
Exp/Cntr=0.3,0.1

Type RM Length L Ch R = 1 ,129297  ,212,202.1,181.8
XS GIS Cut Line= 3
2342282.42641407672388.9215302522342513.24378394672016.062701999
2342515.78023855671785.245332129
#Sta/Elev= 30
       0 2927.53    13.8 2917.99    53.4 2894.08    62.1 2887.08      75 2884.72
    84.4 2877.59      97 2870.12   147.7 2841.26   169.1 2830.95   183.2 2821.11
   192.6 2818.88   227.7 2798.87   239.6  2790.1   244.3 2788.42     249 2788.17
   253.1 2788.24   294.6 2788.21   306.2 2788.62   338.1 2793.91   368.1 2795.74
     409 2803.88   413.7 2803.91   425.3 2801.51   436.9 2804.36   461.4 2805.55
   501.4 2816.89   513.4 2821.53   573.4  2836.8   653.4 2850.41   669.4 2853.96
#Mann= 5 ,-1,0
       0      .1       0   253.1    .045       0   294.6      .1       0
     390     .06       0  598.52      .1       0
Bank Sta=253.1,294.6
XS Rating Curve= 0 ,0
Exp/Cntr(USF)=0,0
Exp/Cntr=0.3,0.1

Type RM Length L Ch R = 1 ,129095  ,250.4,247.5,246.6
XS GIS Cut Line= 3
2342665.43522899 672397.611805112342577.72478685  671972.5283788
2342577.19333542671834.700530645
#Sta/Elev= 30
       0 2933.86     6.2 2933.04    16.8 2928.89    53.5 2906.04      74 2897.58
   102.5 2878.12   118.9 2863.89   127.1 2858.29   151.6 2835.43   158.5 2827.18
   167.9 2811.73   180.1 2803.09   200.6 2792.86   238.4 2789.87   253.7 2788.06
   265.9 2788.28   274.1 2788.55   285.8 2791.84   298.6 2799.46   323.1  2803.6
   339.4 2800.89   351.7 2803.22   407.7 2807.12   433.4 2814.06   441.4 2814.24
   453.4 2817.96   489.4 2825.35   505.4 2831.24   533.4 2835.99   571.9 2845.39
#Mann= 5 ,-1,0
       0      .1       0   238.4    .045       0   265.9      .1       0
     350     .06       0  454.04      .1       0
Bank Sta=238.4,265.9
XS Rating Curve= 0 ,0
Exp/Cntr=0.3,0.1

Type RM Length L Ch R = 1 ,128848  ,190.8,193.5,196.2
XS GIS Cut Line= 2
2342910.27795963672281.8394155732342760.66541038671780.811343679
#Sta/Elev= 30
       0 2902.77     4.9  2901.2    13.2  2900.7    21.5  2896.1    38.3 2881.21
    49.3 2866.16      55 2860.24    84.2 2837.63   100.9 2820.71   108.3 2815.13
   117.6  2810.9   125.9 2804.34   138.4 2797.37   146.9 2794.28   155.1 2789.33
     163 2788.13   196.9 2787.25   201.1 2787.28   233.7 2790.71   242.8 2795.27
   256.2 2799.63   267.9 2797.16   280.4 2799.78   292.9 2798.29   305.4 2799.05
   330.5 2807.54   355.8 2819.31   376.4 2826.48   413.7 2833.67   522.9 2851.75
#Mann= 5 ,-1,0
       0      .1       0     163    .045       0   201.1      .1       0
     240     .06       0     340      .1       0
Bank Sta=163,201.1
XS Rating Curve= 0 ,0
Exp/Cntr(USF)=0,0
Exp/Cntr=0.3,0.1

Type RM Length L Ch R = 1 ,128654  ,255.7,256.8,260.1
XS GIS Cut Line= 2
2343073.51114738672248.9080475092342979.72414738      671641.396
#Sta/Elev= 30
       0  2853.9    28.1 2849.11    71.1 2837.28     105  2824.5   125.2 2814.52
   137.3 2805.53   169.7 2789.56   181.9 2787.89   202.1 2786.59   221.8 2787.45
   254.7 2789.29   266.9 2792.23     283 2793.75   299.2 2793.76   315.4 2790.43
   351.8 2801.06   376.1 2810.49   388.3 2816.95   397.1  2823.4   408.5 2827.33
   428.7  2839.7   452.8 2851.31   465.2 2858.54   493.5 2870.91   509.7  2876.7
   517.8 2877.39   546.1 2888.63   558.3 2890.86   590.6 2904.98   614.7 2912.86
#Mann= 4 ,-1,0
       0      .1       0   181.9    .045       0   221.8     .06       0
     300      .1       0
Bank Sta=181.9,221.8
XS Rating Curve= 0 ,0
Exp/Cntr=0.3,0.1

Type RM Length L Ch R = 1 ,128398  ,361.4,402.8,430.8
XS GIS Cut Line= 3
2343170.88864747672264.5233725422343300.63402136672124.185455299
2343280.06597237671727.783056474
#Sta/Elev= 30
       0  2822.8    13.7 2819.59    64.5 2814.09    79.7 2810.33    99.5 2807.24
   119.7 2801.58   139.1  2797.8   162.5  2796.3   194.1 2796.73   209.7 2795.79
   266.2 2796.72   270.2 2795.93   278.2 2789.95   303.7 2787.42   318.3 2786.05
   345.9 2787.38   370.4 2790.16   402.4 2789.89   411.5 2791.89   442.5 2807.92
   462.5 2821.59   490.5 2837.32   506.6 2848.27   518.6 2857.88   540.9 2871.51
   554.6 2876.13   570.6 2888.39   574.6 2890.73   582.7 2892.96   588.1 2896.15
#Mann= 5 ,-1,0
       0      .1       0   303.7    .045       0   345.9      .1       0
  361.12     .06       0  461.12      .1       0
#XS Ineff= 2 , 0
          262.29 2803.07
Permanent Ineff=
       F       F
Bank Sta=303.7,345.9
XS Rating Curve= 0 ,0
Exp/Cntr(USF)=0,0
Exp/Cntr=0.3,0.1

Type RM Length L Ch R = 1 ,127995  ,175.2,175.2,174.3
XS GIS Cut Line= 3
2343234.50646151 672216.982102152343382.90621734672217.676587097
2343723.30439166672287.965010187
#Sta/Elev= 30
       0 2809.88     9.5  2806.1    21.7 2803.36    61.6 2797.29   101.7 2795.85
   113.7 2796.27   186.5 2792.82     211 2793.89   223.2 2793.46   239.6 2792.34
   243.6 2791.37   255.9 2786.16   264.6  2785.3   268.1 2785.18     298 2785.38
     309 2785.49   313.1 2786.53   321.2  2792.6   325.3 2794.69   333.5 2797.04
   337.6 2799.65     342 2803.89   349.8 2814.33   353.9 2818.79   374.3 2834.96
   390.7 2846.69   439.7 2873.78   451.9 2881.44   488.7 2900.11     496 2902.69
#Mann= 4 ,-1,0
       0      .1       0   264.6    .045       0     298      .1       0
   348.4     .06       0
Bank Sta=264.6,298
XS Rating Curve= 0 ,0
Exp/Cntr=0.3,0.1

Type RM Length L Ch R = 1 ,127820  ,179.4,187.1,189.1
XS GIS Cut Line= 2
2343162.62891714672357.1364716242343692.74793145672453.521746955
#Sta/Elev= 30
       0  2823.6    38.2  2810.7    54.4  2804.1    66.6 2802.41      77 2798.66
    82.9 2797.57   131.7 2797.05   142.4 2797.86   164.2 2796.86   176.4 2794.41
   188.6 2793.35   228.4  2791.7   242.2 2788.78   257.7 2788.18   286.2 2784.49
   290.1 2784.44   321.3 2784.99   330.9  2786.8   341.9 2794.02   355.3 2798.45
   363.4 2804.65   375.6  2811.3   391.9 2822.06     400 2826.48   444.7 2852.73
     461 2858.53   505.7 2881.06   513.7 2886.01   530.1 2899.19   538.8 2902.48
#Mann= 5 ,-1,0
       0      .1       0   286.2    .045       0   321.3      .1       0
     400     .06       0     500      .1       0
Bank Sta=286.2,321.3
XS Rating Curve= 0 ,0
Exp/Cntr(USF)=0,0
Exp/Cntr=0.3,0.1

Type RM Length L Ch R = 1 ,127633  ,287.1,277.5,272.9
XS GIS Cut Line= 2
2343068.12612912672426.7619208192343573.46026066  672669.0373106
#Sta/Elev= 30
       0 2858.62     4.8 2853.99     8.9 2851.44    22.2 2849.91    26.7  2847.9
    37.8 2839.31    61.8 2827.22    67.8 2823.16    79.9 2820.43    97.6 2810.18
   124.3 2802.03     142 2799.13   186.4 2798.21   204.1 2796.04   226.3 2791.76
   256.7 2791.49   274.7 2787.54   329.4 2785.02   346.7 2784.57   354.9 2785.11
   361.7 2787.17   377.1 2788.71   409.6 2787.06   421.5 2791.04   439.2 2794.06
   477.5 2806.63   510.2 2822.31   536.8 2830.86   545.7 2834.63   560.4 2838.64
#Mann= 5 ,-1,0
       0      .1       0     320     .06       0   329.4    .045       0
   354.9     .06       0     520      .1       0
Bank Sta=329.4,354.9
XS Rating Curve= 0 ,0
Exp/Cntr=0.3,0.1

Type RM Length L Ch R = 1 ,127355  ,226.7,219.5,217.1
XS GIS Cut Line= 2
2342861.38354666 672803.521787982343587.31685717672835.481116116
#Sta/Elev= 30
       0 2915.11    66.9 2918.55   130.9 2914.53   162.9 2907.04     195 2902.03
     203 2898.79   256.7 2862.38     259 2860.56     267 2848.75   271.1 2844.11
   284.2  2833.6   319.5 2813.24   347.1 2799.07   363.1 2789.23   383.2 2784.03
   406.9 2783.72   418.4  2783.8   427.2 2784.54   435.2 2786.85   467.2 2788.59
   503.3 2788.39   531.3  2792.5   547.3 2792.07   566.6 2794.46   591.4  2800.9
   627.4 2814.81   635.4 2816.76   663.4 2828.45   691.5 2834.89   726.6 2844.78
#Mann= 5 ,-1,0
       0      .1       0   383.2    .045       0   418.4      .1       0
     600     .06       0     700      .1       0
Bank Sta=383.2,418.4
XS Rating Curve= 0 ,0
Exp/Cntr(USF)=0,0
Exp/Cntr=0.3,0.1

Type RM Length L Ch R = 1 ,127136  ,160.2,164.1,166.7
XS GIS Cut Line= 3
     2342891.017673136.894511862 2343394.4291469673014.034127965
2343604.61774886672979.784317517
#Sta/Elev= 30
       0 2816.76    34.1 2820.96    46.5 2820.69    54.7 2822.76    71.2 2822.47
   137.1 2826.88   165.9 2826.72   207.1 2828.72   305.9 2827.33   322.3 2825.24
   338.8 2820.82   354.9 2814.54   371.8 2802.67   383.2 2792.83   396.5 2784.42
   425.3 2783.27     454 2783.22   464.1 2783.49   507.6 2790.66     520 2791.97
   536.2 2791.58   560.5 2794.75   568.6 2794.17   584.8  2797.9     597 2797.41
     623 2801.62   665.9 2815.53     678 2821.25   718.5 2833.93   731.1 2836.21
#Mann= 5 ,-1,0
       0      .1       0   425.3    .045       0   464.1      .1       0
  588.19     .06       0  678.19      .1       0
Bank Sta=425.3,464.1
XS Rating Curve= 0 ,0
Exp/Cntr=0.3,0.1

Type RM Length L Ch R = 1 ,126972  ,308.6,309.7,311.9
XS GIS Cut Line= 2
2342900.37869475673251.4285303712343686.67962508673144.897436585
#Sta/Elev= 30
       0 2801.31      20 2797.61    44.2 2802.31    56.3 2802.83    72.5 2805.51
     129 2807.12   161.3 2809.07   193.8 2808.13   221.3 2809.04   258.1 2811.86
   286.4 2811.63   306.6 2808.59   338.9 2795.99   346.9 2794.79   367.1 2789.58
   403.4 2787.47   445.4 2783.32   463.7 2782.38   500.3 2783.03   520.5 2789.68
     577 2794.03   629.5 2805.99   665.8 2817.26   677.3 2819.67   698.1    2828
   706.2 2829.67   726.4 2837.27   738.5 2839.29   746.6 2842.34   793.5 2854.82
#Mann= 5 ,-1,0
       0     .12       0      70      .1       0   445.4    .045       0
   500.3     .06       0     560      .1       0
Bank Sta=445.4,500.3
XS Rating Curve= 0 ,0
Exp/Cntr(USF)=0,0
Exp/Cntr=0.3,0.1
