HEC-RAS study GLADYFK.prj: GLADYFK

--- GLADYFK.g01 (geometry) --- (continued)

Type RM Length L Ch R = 1 ,70292   ,511.8,491.1,464.8
XS GIS Cut Line= 4
2355526.31464466698671.1098069432355828.47241882 698829.74263838
2356012.78279589698924.3286112812356118.93821788 698903.74994012
#Sta/Elev= 30
       0 2581.88    13.1  2581.2      71 2585.66    91.8 2586.08   119.6    2582
   169.3 2580.41   176.6 2578.42   187.3 2572.02   198.4  2571.3   242.9 2571.15
   245.8 2571.19   264.1 2572.94   278.4 2572.11   291.2 2574.87   318.3 2574.56
   331.9 2575.58   367.9 2573.34   381.4 2575.48   394.9 2575.95   417.9 2574.27
   466.8 2573.78   480.3 2572.22   507.3 2579.12   564.3 2578.07   592.6 2581.49
   600.8 2581.57   604.9 2582.17     613 2585.71   637.5 2593.41   656.6 2597.19
#Mann= 5 ,-1,0
       0      .1       0   198.4    .045       0   245.8      .1       0
  491.27     .06       0  598.43      .1       0
#XS Ineff= 2 , 0
                          526.29         2582.85
Permanent Ineff=
       F       F
Bank Sta=198.4,245.8
XS Rating Curve= 0 ,0
Exp/Cntr(USF)=0,0
Exp/Cntr=0.3,0.1

Type RM Length L Ch R = 1 ,69801   ,195,193,189.7
XS GIS Cut Line= 2
2355541.42253337699348.4468173652356163.36395186698910.318044824
#Sta/Elev= 30
       0 2706.27    18.7 2694.63    27.3 2688.11    32.7 2681.95    47.4 2673.56
    70.3 2656.16      96 2640.57   110.5 2628.23   130.6 2614.88   174.6 2579.56
   202.4 2570.32   227.9 2569.53   241.8 2570.62   274.2 2573.56   359.9 2570.61
   394.8 2572.65   411.7 2570.55   443.7 2573.37   468.2 2572.65   482.9 2569.97
   497.5 2572.83   536.7 2573.73   549.7 2577.85   561.2 2578.97     615 2577.29
   635.9 2580.54   649.2 2580.55   668.8 2591.78   693.3 2593.57   760.8 2609.06
#Mann= 5 ,-1,0
       0      .1       0   202.4    .045       0   241.8      .1       0
     630     .06       0     730      .1       0
#XS Ineff= 2 , 0
                           576.6         2586.53
Permanent Ineff=
       F       F
Bank Sta=202.4,241.8
XS Rating Curve= 0 ,0
Exp/Cntr(USF)=0,0
Exp/Cntr=0.3,0.1

Type RM Length L Ch R = 1 ,69608   ,470.4,468.3,448.7
XS GIS Cut Line= 3
 2355731.4265376 699475.802682452355962.98902866699255.835767545
2356170.15810441699043.036386382
#Sta/Elev= 30
       0 2667.98    21.2 2650.28    50.7 2631.54    67.5 2618.78    83.8 2604.46
    92.9  2599.2     120 2579.93   137.4 2569.72     149 2568.96   163.7 2568.95
   183.9    2569   194.8 2569.16   218.7 2571.98   236.1  2571.4   248.5  2569.7
   271.2 2572.38   288.4 2572.76     344 2571.02   406.8 2572.93   423.6  2571.5
   435.2 2571.92   446.6 2569.12     453 2569.04   475.9 2573.85   497.5  2575.8
   521.8 2576.12   534.3 2578.41   545.6 2578.79   568.7 2587.85   616.4 2598.58
#Mann= 4 ,-1,0
       0      .1       0     149    .045       0   183.9      .1       0
  499.38     .06       0
Bank Sta=149,183.9
XS Rating Curve= 0 ,0
Exp/Cntr(USF)=0,0
Exp/Cntr=0.3,0.1

Type RM Length L Ch R = 1 ,69139   ,238.4,234.1,231.6
XS GIS Cut Line= 2
2356078.55621811699622.2321100922356266.60848319699096.453328139
#Sta/Elev= 30
       0 2649.66    13.9 2641.14    52.1    2614    60.6  2606.7    77.6 2589.09
    86.1 2582.18    94.6 2573.06    98.8 2569.95   103.1 2568.58   115.8 2568.43
   124.3  2570.4   152.3 2572.34   200.8 2572.91     222 2570.21   247.5 2571.18
   260.3 2567.86     273 2569.36   302.5 2569.82   325.5  2567.5   346.3 2570.78
   370.7 2569.97   390.1 2567.31   413.2 2566.99   417.4    2567   425.9 2568.05
   434.4 2575.96     437 2576.85   451.4 2578.91   468.4 2585.89   558.4 2608.46
#Mann= 5 ,-1,0
       0      .1       0     320     .06       0   390.1    .045       0
   417.4     .06       0     510      .1       0
Bank Sta=390.1,417.4
XS Rating Curve= 0 ,0
Exp/Cntr(USF)=0,0
Exp/Cntr=0.3,0.1

Type RM Length L Ch R = 1 ,68905   ,237.1,217.3,212.4
XS GIS Cut Line= 2
2356354.87791373699599.2053021242356462.33635092699207.749566655
#Sta/Elev= 30
       0 2607.74     2.1 2605.78    10.4  2600.7    22.8 2588.93    39.4 2574.91
    51.9 2568.37      56 2566.92    64.3  2566.1    84.1 2567.09    95.6 2566.64
   110.1 2568.12   126.5 2566.42   130.7 2566.96   139.4 2569.76   159.7 2570.42
   192.9 2569.02   213.6  2569.3     224 2566.73   235.5 2566.14   242.7 2566.03
   286.9 2566.12   300.8 2566.97   304.9 2568.49   313.2 2573.29   315.1 2573.76
   321.5 2574.82   338.1 2575.43   350.5 2581.32   373.7 2586.84   405.9 2592.94
#Mann= 5 ,-1,0
       0      .1       0   235.5    .045       0   286.9      .1       0
     290     .06       0     390      .1       0
Bank Sta=235.5,286.9
XS Rating Curve= 0 ,0
Exp/Cntr(USF)=0,0
Exp/Cntr=0.3,0.1

Type RM Length L Ch R = 1 ,68688   ,236.9,235.6,234.7
XS GIS Cut Line= 2
2356727.14464256699568.5028914992356558.28138413699188.560560014
#Sta/Elev= 30
       0 2638.05    12.4 2628.74    16.8 2624.73    35.1 2605.56      43 2594.26
    50.2 2587.08    69.3 2572.37    74.5 2569.46    82.4 2566.31    95.6 2564.72
   115.6 2564.83   117.4    2565   126.2 2568.76   139.3 2569.45   162.3 2568.93
   177.5 2567.81   192.7 2564.67   200.6 2564.29   226.9 2564.43     240 2566.09
   253.1 2565.82   286.6 2568.03     329 2568.03   332.1 2568.52   345.1 2572.99
   358.2 2573.66   371.3 2579.19   389.6 2584.04   398.7 2587.19   415.8 2591.44
#Mann= 4 ,-1,0
       0      .1       0   192.7    .045       0   226.9      .1       0
     270     .06       0
Bank Sta=192.7,226.9
XS Rating Curve= 0 ,0
Exp/Cntr(USF)=0,0
Exp/Cntr=0.3,0.1

Type RM Length L Ch R = 1 ,68452   ,337.7,317.2,303.3
XS GIS Cut Line= 3
2356945.89931827699445.6932489992356803.90066913699180.884957358
2356669.57762264699061.913116186
#Sta/Elev= 30
       0 2644.35    28.2 2625.33      46 2611.28    50.5 2606.84    59.6 2596.15
    73.2 2583.05    82.3 2575.76    93.2 2565.61    95.9  2563.8   100.4 2562.83
   145.8 2566.82     164 2566.59   178.9 2564.52   191.2  2563.7   232.1 2563.56
     238 2563.93   250.2 2567.97   258.7 2569.84   268.4  2569.2   321.5 2568.67
   339.7  2570.2   353.5 2572.97   362.4 2572.84   368.1 2574.85   376.6 2579.14
   393.6 2584.73   421.9 2596.06   438.8 2601.77   460.4 2611.04   479.9 2616.75
#Mann= 5 ,-1,0
       0      .1       0   191.2    .045       0   232.1      .1       0
     260     .06       0  390.48      .1       0
Bank Sta=191.2,232.1
XS Rating Curve= 0 ,0
Exp/Cntr(USF)=0,0
Exp/Cntr=0.3,0.1

Type RM Length L Ch R = 1 ,68135   ,311.6,309.4,312.6
XS GIS Cut Line= 2
2357270.96768194699184.3975085512356761.77587733698929.801606244
#Sta/Elev= 30
       0  2674.1    34.3 2655.31    56.8 2640.34    67.1 2636.36    79.1 2626.05
     106 2606.01   126.7 2588.95   141.4 2574.26   150.3 2563.51   153.6 2562.26
   195.3 2561.63   208.8 2562.42   228.1 2565.05   248.7 2563.96   271.5 2567.77
   314.5 2567.35   338.5 2569.41   359.3 2569.49   371.2 2567.95   401.1 2568.09
     410 2568.79   423.5 2572.46   436.8 2573.25   478.5 2597.74   495.1 2605.93
   508.3 2615.87   517.4 2620.65   547.1 2631.86   553.2 2635.13   569.3  2638.4
#Mann= 5 ,-1,0
       0      .1       0   153.6    .045       0   208.8      .1       0
     380     .06       0     490      .1       0
Bank Sta=153.6,208.8
XS Rating Curve= 0 ,0
Exp/Cntr(USF)=0,0
Exp/Cntr=0.3,0.1

Type RM Length L Ch R = 1 ,67826   ,284,285.1,286.2
XS GIS Cut Line= 2
2357430.43984053 698921.408334742356868.09064972698633.239346415
#Sta/Elev= 30
       0 2668.74    10.8 2664.91      34 2653.64    74.5 2631.24    85.1 2627.18
   108.8 2613.49   119.4  2610.1   128.4 2605.42   146.4 2589.32   162.3 2570.58
   173.3 2563.63   218.8 2562.33   245.3 2560.94   276.7 2562.06   287.1 2561.38
   303.7 2565.43   326.2 2563.67   358.5 2566.41   384.6 2565.71   400.1 2569.63
     416 2569.84   429.5 2577.92   474.4 2597.11     488 2605.44     516 2615.77
   553.1 2636.07   563.5 2639.93   575.4 2647.92   609.3 2660.32   631.9 2666.83
#Mann= 5 ,-1,0
       0      .1       0   218.8    .045       0   276.7      .1       0
     420     .06       0     560      .1       0
Bank Sta=218.8,276.7
XS Rating Curve= 0 ,0
Exp/Cntr(USF)=0,0
Exp/Cntr=0.3,0.1

Type RM Length L Ch R = 1 ,67541   ,200.1,200.9,201.6
XS GIS Cut Line= 2
2357553.54115593698675.2057039382357058.33813716698395.429987117
#Sta/Elev= 30
       0 2648.45    90.6 2606.27   122.9 2590.48   162.4 2577.74   181.6 2565.57
   212.9  2559.7   228.5 2559.34   263.8 2559.54   295.6 2560.33   304.8 2563.12
     314 2563.64   328.3 2562.81   359.9 2564.21   369.1 2562.86   381.2 2563.17
   401.3 2567.08   410.5    2571     427 2580.37   448.7 2590.61   457.5 2596.33
   469.3 2598.75   472.2 2600.07   483.9 2608.33   506.9 2619.56   516.4 2622.62
   529.9 2631.02     549 2636.48   552.9 2637.97   562.1 2643.39   568.8 2645.88
#Mann= 5 ,-1,0
       0      .1       0   212.9    .045       0   263.8      .1       0
     290     .06       0     490      .1       0
Bank Sta=212.9,263.8
XS Rating Curve= 0 ,0
Exp/Cntr(USF)=0,0
Exp/Cntr=0.3,0.1

Type RM Length L Ch R = 1 ,67340   ,307.6,319,317.4
XS GIS Cut Line= 2
2357643.06938531698504.5425166772357181.43945256698221.969042689
#Sta/Elev= 30
       0 2645.91    40.9 2625.81    50.3 2622.36    59.8 2616.36    83.1 2607.58
   111.3 2592.75     129 2586.11   139.4  2578.5   148.8 2573.97   167.5 2567.94
   179.1 2560.02   211.1 2558.91   237.9 2558.29   248.9 2558.79   284.8 2561.58
   335.9 2559.34   345.8 2561.58   383.3 2561.17     402 2565.76   406.7 2567.88
   432.2 2585.18   443.2 2589.88   448.9 2597.15   453.6 2601.01     463 2604.09
   472.9 2610.54   486.5 2615.06   500.5 2622.92   509.9 2625.28   541.2 2637.39
#Mann= 5 ,-1,0
       0      .1       0   211.1    .045       0   248.9      .1       0
     320     .06       0     490      .1       0
Bank Sta=211.1,248.9
XS Rating Curve= 0 ,0
Exp/Cntr(USF)=0,0
Exp/Cntr=0.3,0.1

Type RM Length L Ch R = 1 ,67021   ,400,441.3,479.3
XS GIS Cut Line= 3
  2357766.746688698346.7912376172357684.17707366698180.936451278
2357408.48711777 697981.93791351
#Sta/Elev= 30
       0 2640.64     6.3 2638.87    19.7  2632.3    46.5 2624.82    65.8 2615.94
    73.3 2611.52    86.6 2608.99    95.6 2601.87   104.6 2599.11   153.7  2570.9
   164.2 2566.63   176.1 2563.64   212.2 2564.04   222.3 2559.38   230.9 2557.72
     279 2558.01   331.2 2556.37   343.1 2556.48   368.5 2556.72   376.2 2557.95
   388.5 2561.79   403.6 2558.41   422.1 2557.96   436.9 2559.17   451.7 2568.17
   461.5 2577.35   471.9 2584.27   500.3 2596.13   515.8 2609.65   525.3 2615.76
#Mann= 5 ,-1,0
       0      .1       0     279    .045       0   343.1      .1       0
  385.27     .06       0  505.27      .1       0
Bank Sta=279,343.1
XS Rating Curve= 0 ,0
Exp/Cntr(USF)=0,0
Exp/Cntr=0.3,0.1

Type RM Length L Ch R = 1 ,66580   ,285.1,289.5,299.5
XS GIS Cut Line= 6
2357876.70765945698282.5087722052357833.01416437698103.937993868
 2357823.1765303698010.9276353552357840.24611279697956.175651552
2357902.77546907697796.5344857562357937.68965532697688.618847806
#Sta/Elev= 30
       0 2632.03    34.3 2619.97    46.7 2613.92      59 2612.77   104.3 2595.81
   124.9 2585.34   137.3 2581.33     162 2569.83   170.3 2568.44   178.4 2564.31
   186.6 2562.29   234.4 2560.23   246.9 2563.23     259 2562.26   270.8 2562.87
   304.3 2558.98   333.7 2559.14   346.5 2556.58   364.8 2558.06   395.6 2554.24
   449.6 2554.17   453.1 2554.19   462.5 2554.24   471.1 2557.93   488.3 2570.43
   506.2 2588.69   525.8  2602.5   551.2 2623.72   602.4 2659.28   619.6 2669.57
#Mann= 5 ,-1,0
       0      .1       0  354.72     .06       0   395.6    .045       0
   453.1     .06       0  454.72      .1       0
#XS Ineff= 2 , 0
           248.9 2585.73
Permanent Ineff=
       F       F
Bank Sta=395.6,453.1
XS Rating Curve= 0 ,0
Exp/Cntr=0.3,0.1

Type RM Length L Ch R = 1 ,66290   ,230.5,233.2,246.2
XS GIS Cut Line= 4
2357986.90854899698276.5089325772358042.28747103698122.718931644
2358074.79608498 698078.549550092358242.04041298697862.355662674
#Sta/Elev= 30
       0  2594.9     3.7 2593.31      38  2585.1    54.6 2579.35    63.1 2578.74
    71.6  2575.9    84.3 2575.48    98.2 2572.39   126.8 2568.89   144.3 2563.89
   156.8 2563.56   171.6 2561.13   190.2 2560.31   205.1 2557.38   235.2 2557.47
   251.6  2555.9   270.6 2552.26   285.9 2552.12   322.9 2552.26   336.3 2552.39
   342.9 2554.26   351.3 2560.79   376.8 2583.54   399.9 2597.33   414.2 2608.11
     437 2622.62   442.8 2627.28   454.1 2631.65   462.6 2637.73   491.6 2652.29
#Mann= 5 ,-1,0
       0      .1       0   268.3     .06       0   270.6    .045       0
   322.9     .06       0   388.3      .1       0
Bank Sta=270.6,322.9
XS Rating Curve= 0 ,0
Exp/Cntr(USF)=0,0
Exp/Cntr=0.3,0.1

Type RM Length L Ch R = 1 ,66057   ,248.6,252.1,258.2
XS GIS Cut Line= 4
2357985.28384708698345.6125298852358157.27855801698286.128432286
2358195.85017512698256.8865538542358499.30018068698037.547683805
#Sta/Elev= 30
       0 2611.17    28.5 2597.67    43.5 2591.92    70.8 2582.92   100.4 2575.28
   113.1 2573.55   144.1 2567.29   155.4 2563.53   168.1 2562.47   176.6 2560.29
   190.4 2558.36     199 2558.78   216.7 2556.19   240.7 2556.09   277.7 2550.91
   280.1 2550.85   314.7 2550.98   344.3 2552.83   382.3 2566.84   413.4 2581.71
   441.6 2593.18   456.7 2600.73   462.8 2602.94   475.7 2611.76   487.4 2617.83
   507.2 2631.51   519.8 2638.66   536.8 2650.93   553.6 2661.19   604.8  2683.4
#Mann= 5 ,-1,0
       0      .1       0   277.7    .045       0   314.7      .1       0
  380.39     .06       0  500.39      .1       0
Bank Sta=277.7,314.7
XS Rating Curve= 0 ,0
Exp/Cntr=0.3,0.1

Type RM Length L Ch R = 1 ,65805   ,215.8,214.6,213.4
XS GIS Cut Line= 2
2358099.41248235 698549.984588072358549.33896707698369.725570946
#Sta/Elev= 30
       0 2616.68    22.4 2601.73      35 2594.87    48.2 2589.95    61.1 2582.76
   112.9 2561.22   130.1 2560.55   138.7 2557.68   147.3 2556.41   177.5 2557.08
   194.7 2555.19   207.3 2554.71   224.9 2555.47   238.1 2550.31   253.5 2549.87
   276.6 2549.77   302.5  2549.8   336.9  2550.7   341.2 2551.59   349.9 2557.63
   370.4 2566.93   379.6 2573.37   384.3 2575.78   401.6 2581.78   410.2 2586.95
   418.8 2590.55     436 2602.61   453.5 2610.65   479.1 2626.72   484.7 2629.57
#Mann= 4 ,-1,0
       0      .1       0   253.5    .045       0   302.5      .1       0
     340     .06       0
Bank Sta=253.5,302.5
XS Rating Curve= 0 ,0
Exp/Cntr(USF)=0,0
Exp/Cntr=0.3,0.1

Type RM Length L Ch R = 1 ,65590   ,262.9,264.3,266.7
XS GIS Cut Line= 3
2358147.26071094698779.6703943872358575.12024322698581.937655317
  2358751.731836698501.097904098
#Sta/Elev= 30
       0 2647.61      25 2628.09    45.9 2614.19    62.7 2604.55    75.9 2594.32
     108    2576     142 2560.64   155.2 2559.71     164  2556.2     177 2554.71
   213.5 2555.92     239  2555.1   269.8 2553.21     283 2549.27   294.9 2549.02
   313.9 2548.73   340.9 2548.99   358.7 2549.68   364.2    2551     380 2562.74
     424 2585.52   485.7 2606.97   525.3 2626.06   534.1 2628.04   554.2 2638.62
   598.1 2657.94   608.9 2660.94   626.6 2668.41   635.3 2668.99   665.6 2680.84
#Mann= 6 ,-1,0
       0      .1       0   294.9    .045       0   340.9      .1       0
     350     .08       0     410     .06       0  511.34      .1       0
Bank Sta=294.9,340.9
XS Rating Curve= 0 ,0
Exp/Cntr=0.3,0.1

Type RM Length L Ch R = 1 ,65326   ,192.2,197.8,198.7
XS GIS Cut Line= 2
2358268.58460041698981.4883726982358713.11712825698826.057418909
#Sta/Elev= 30
       0 2634.76    16.5 2620.94    34.5 2607.33    53.3 2589.65    63.1 2581.77
    67.4 2578.61    75.8 2575.47      97 2560.64   101.3 2559.06   109.8 2558.02
   122.4 2554.32   139.4  2553.7   152.1 2553.98   160.6 2552.95   177.5 2552.35
   188.3 2550.06   194.5 2548.07     204 2547.94   244.8 2547.67   254.2 2547.85
   287.7 2550.06   296.2 2549.73   304.7 2552.21   313.1  2553.8     347 2569.06
     364 2577.57   379.8 2584.19   440.3 2607.72   457.2 2616.78   470.9 2623.44
#Mann= 6 ,-1,0
       0      .1       0     204    .045       0   254.2      .1       0
     260     .08       0     370     .06       0     470      .1       0
Bank Sta=204,254.2
XS Rating Curve= 0 ,0
Exp/Cntr(USF)=0,0
Exp/Cntr=0.3,0.1

Type RM Length L Ch R = 1 ,65128   ,286.2,285.3,279.6
XS GIS Cut Line= 4
2358297.82505975699178.3006394672358435.06945849699115.818528709
2358661.33504218699068.4190190832358809.57512077699003.081426261
#Sta/Elev= 30
       0 2651.96    33.3 2640.23    46.5 2631.72    59.7 2627.39    64.1 2624.21
    72.9  2615.2    93.2  2600.7   103.7 2590.97   114.4  2585.2   151.9 2558.39
   160.1 2556.91   174.2 2550.95   209.1 2546.97   262.6    2547   270.4 2546.83
   290.9  2548.2   299.1 2551.62   303.1 2551.88   315.4 2552.28   348.1 2549.71
   353.3 2550.84   360.4 2554.02   376.7 2567.52   380.8 2569.83     420  2584.9
   449.5 2594.42   481.2 2607.03   499.1 2614.78     514 2623.65     544  2636.5
#Mann= 5 ,-1,0
       0      .1       0   209.1    .045       0   262.6     .08       0
   330.8     .06       0  481.98      .1       0
Bank Sta=209.1,262.6
XS Rating Curve= 0 ,0
Exp/Cntr=0.3,0.1

Type RM Length L Ch R = 1 ,64843   ,203.1,205.7,219
XS GIS Cut Line= 2
2358389.82074437699435.3467577622358856.11360573699283.024423049
#Sta/Elev= 30
       0 2603.78    19.3 2599.88    31.9 2595.06    54.3 2588.77    73.4 2579.65
    90.8 2574.03     110 2566.09   114.6 2562.85   120.9 2556.54   124.5 2554.68
   132.9 2554.23   141.3 2548.41     154 2545.84   162.4 2545.75   212.8 2545.53
   222.4 2545.74   241.5 2546.41     251  2549.6   279.5 2550.79   318.1 2549.73
   334.9 2547.19   355.9 2548.68   360.2 2550.42   371.5 2560.58   381.2 2566.74
   389.6 2570.71   402.2  2574.8   425.3 2585.16   440.1 2593.38   490.5 2618.48
#Mann= 4 ,-1,0
       0      .1       0   162.4    .045       0   222.4      .1       0
     440     .06       0
Bank Sta=162.4,222.4
XS Rating Curve= 0 ,0
Exp/Cntr(USF)=0,0
Exp/Cntr=0.3,0.1

Type RM Length L Ch R = 1 ,64637   ,280.4,286.5,303.8
XS GIS Cut Line= 3
2358374.61720078699603.9681854862358709.85907257699572.483148389
2358996.63829678699542.199055646
#Sta/Elev= 30
       0 2594.02     5.6 2593.03    29.7 2584.88    57.8 2578.42    77.9  2574.5
      94 2572.81     145 2562.46   154.6 2559.21   165.6 2554.27   178.3  2553.1
   182.4 2551.99   190.4 2547.46   194.4 2546.25     206 2546.04   262.7 2544.89
   286.8 2545.37   286.8 2545.38   302.9 2546.75   314.9 2546.33     323 2547.93
     339  2548.4   395.4 2544.63   411.4 2546.82   415.5 2548.35     448 2571.62
   479.8 2590.64     520 2609.38   589.2 2633.99   608.5 2639.17   625.1  2644.8
#Mann= 4 ,-1,0
       0      .1       0     206    .045       0   286.8      .1       0
  536.72     .06       0
Bank Sta=206,286.8
XS Rating Curve= 0 ,0
Exp/Cntr=0.3,0.1

Type RM Length L Ch R = 1 ,64351   ,206.9,208.2,214.8
XS GIS Cut Line= 2
2358430.95498783699802.4947380252358942.10522246700001.415272684
#Sta/Elev= 30
       0 2567.65    24.6 2565.18    48.5 2561.09    65.7 2555.06    78.6 2554.88
    95.7 2553.28   112.9 2555.21   125.8 2554.78   130.1 2553.77   138.7 2547.79
     143 2545.82   151.3 2543.76   172.8 2543.34   185.9 2544.35   241.7  2548.1
   254.6 2545.97   280.3 2545.18   301.8 2547.73   358.3 2544.45   374.7 2546.19
     380 2547.96   421.9 2574.15   460.6 2596.69   469.2 2602.94   477.7  2611.6
   486.3 2616.63   499.2 2620.27   520.7 2622.99   542.1 2624.42   548.5 2623.21
#Mann= 3 ,-1,0
       0      .1       0   151.3    .045       0   185.9      .1       0
Bank Sta=151.3,185.9
XS Rating Curve= 0 ,0
Exp/Cntr(USF)=0,0
Exp/Cntr=0.3,0.1

Type RM Length L Ch R = 1 ,64142   ,279.3,291.7,311.9
XS GIS Cut Line= 3
2358285.24788708699931.4826475762358611.74442499700100.397814514
 2358867.0024097700223.405531408
#Sta/Elev= 30
       0 2567.97    57.3 2564.66      82 2561.03    95.4 2556.45   115.9 2553.43
   151.9 2552.87   184.5 2554.39   190.4  2552.7     197  2548.1   210.5 2545.22
   234.9 2546.81   246.5 2543.53   255.5 2544.28   273.5 2542.13   273.5 2542.12
   317.1 2541.74   323.1 2541.91   341.1  2544.1   434.4 2542.43   449.4 2544.93
   470.8 2555.98   501.3 2578.03     519 2593.08   554.6  2613.6   576.8 2622.01
   585.7 2621.12   603.4 2614.95   629.2 2598.31   638.9 2596.67     651 2589.74
#Mann= 3 ,-1,0
       0      .1       0   273.5    .045       0   323.1      .1       0
Bank Sta=273.5,323.1
XS Rating Curve= 0 ,0
Exp/Cntr=0.3,0.1

Type RM Length L Ch R = 1 ,63851   ,292.8,297.4,302.1
XS GIS Cut Line= 3
2358238.22248603700004.0706177892358307.91430599700196.540017919
2358451.94113435700458.786910856
#Sta/Elev= 30
       0 2562.47    55.5 2555.23    77.8 2553.86    94.8    2554   111.5 2551.56
   154.3 2552.52   158.6  2553.4   192.6 2550.81   232.8 2549.79   238.5    2549
   241.9 2547.35   246.6  2543.8   251.1 2542.37   270.2 2540.66     282 2540.68
   343.8 2540.76   379.2 2542.35   385.1 2543.88   396.4 2551.39   401.7 2555.74
   404.7  2559.4   411.6 2570.57   415.4  2575.5   423.3 2582.89   438.1 2594.84
   456.4 2611.48   465.5 2618.86   476.4 2623.59   492.9 2627.35   503.9 2628.95
#Mann= 3 ,-1,0
       0      .1       0     282    .045       0   343.8      .1       0
Bank Sta=282,343.8
XS Rating Curve= 0 ,0
Exp/Cntr(USF)=0,0
Exp/Cntr=0.3,0.1

Type RM Length L Ch R = 1 ,63553   ,325.3,325,327.7
XS GIS Cut Line= 2
 2357962.6674027700028.1798596312358149.18454725700584.277272076
#Sta/Elev= 30
       0 2588.84    34.8 2582.28    74.6 2572.58    98.1 2567.95   161.4 2561.53
   182.5 2560.93   207.8 2556.47   220.4 2551.37   231.2 2550.57   241.5 2548.21
   254.2 2547.76   279.5 2549.04   287.9 2548.69   330.1 2543.48   342.8 2543.91
   365.3 2542.11   380.8 2539.94   387.4 2539.98   432.4 2540.46   456.7 2541.15
   465.1 2549.73   472.7 2555.23     482 2561.27   490.5 2565.39   511.6 2581.26
   532.6 2593.46   545.1 2599.99     558 2605.05   570.5  2612.1   586.5 2616.05
#Mann= 3 ,-1,0
       0      .1       0   387.4    .045       0   432.4      .1       0
#XS Ineff= 2 , 0
          280.84 2558.82
Permanent Ineff=
       F       F
Bank Sta=387.4,432.4
XS Rating Curve= 0 ,0
Exp/Cntr(USF)=0,0
Exp/Cntr=0.3,0.1

Type RM Length L Ch R = 1 ,63228   ,271.2,270.4,269.9
XS GIS Cut Line= 2
2357696.70777067700135.2545166862357814.14449131700649.903674787
#Sta/Elev= 30
       0 2577.88    30.7 2570.27      58 2565.92      68 2563.38   118.1 2557.14
   137.4 2553.11   153.8  2547.7   166.1 2547.55   178.4 2543.66   211.2 2543.17
   223.5 2545.09   228.3 2544.67   239.9 2541.88   267.3 2543.88   289.2 2544.14
   315.2 2542.46   331.9 2539.89   350.7 2539.01     363 2540.45   371.2 2538.87
   388.7 2538.32     412 2538.01   418.7 2538.56   432.8 2540.93     441 2540.56
   445.1 2543.56   453.3 2547.54   483.1 2564.35   514.8 2585.37   527.9 2591.53
#Mann= 3 ,-1,0
       0      .1       0   388.7    .045       0   418.7      .1       0
Bank Sta=388.7,418.7
XS Rating Curve= 0 ,0
Exp/Cntr(USF)=0,0
Exp/Cntr=0.3,0.1

Type RM Length L Ch R = 1 ,62958   ,269.1,266.5,265.3
XS GIS Cut Line= 2
2357430.74813863700207.7889617872357572.36300763700791.518543794
#Sta/Elev= 30
       0 2567.73    71.4 2557.23    79.6 2556.87     129    2545   137.3 2543.72
   149.6 2544.33   161.3 2543.26   174.3 2543.68   182.5 2541.47   207.2  2540.5
   240.8 2540.16   252.5 2541.49   267.3 2539.19   285.4 2542.26   301.9 2541.75
   310.1 2542.78   334.8  2541.6   347.2 2538.33   362.3 2536.53   388.3 2536.44
   409.8 2536.55   433.6 2536.62     446 2540.73   450.1 2543.99   459.4 2553.57
   503.6 2576.92   512.4 2582.77   520.1 2586.27   540.6 2589.94   600.7 2595.21
#Mann= 3 ,-1,0
       0      .1       0   362.3    .045       0   409.8      .1       0
Bank Sta=362.3,409.8
XS Rating Curve= 0 ,0
Exp/Cntr(USF)=0,0
Exp/Cntr=0.3,0.1

Type RM Length L Ch R = 1 ,62691   ,209.1,211.6,209.3
XS GIS Cut Line= 2
2357144.06437942700297.5935128652357340.94358755700877.869073677
#Sta/Elev= 30
       0 2576.16    34.5 2565.43    54.5 2558.04      66 2556.53    79.8 2551.42
   100.9 2546.47   113.6 2545.05   122.1 2543.12   130.5    2543   143.2 2539.61
   244.6 2538.92   261.5 2542.56   280.5  2538.8   307.9 2539.74   324.8 2538.37
   333.3 2535.41   345.9  2535.2   383.9 2535.04   389.1 2535.16   413.5 2535.32
   417.7 2536.68   426.2 2542.73   447.3 2546.04   457.1 2551.44   489.5 2565.58
   519.1 2572.87   544.5 2578.04   564.3 2579.38   583.2 2581.85   612.8 2582.54
#Mann= 5 ,-1,0
       0      .1       0      20     .12       0     220      .1       0
   345.9    .045       0   389.1      .1       0
Bank Sta=345.9,389.1
XS Rating Curve= 0 ,0
Exp/Cntr(USF)=0,0
Exp/Cntr=0.3,0.1

Type RM Length L Ch R = 1 ,62480   ,224.5,203.1,185.7
XS GIS Cut Line= 4
 2356860.8346414700373.5819791622357019.71961638700563.553144904
2357071.52993431700722.4381198882357199.32871854700943.495476388
#Sta/Elev= 30
       0 2618.69    15.1 2611.85    27.6 2604.28    36.2 2601.09    72.5  2580.9
     105 2565.04   117.4 2555.35   124.2 2553.87   129.9 2551.03   144.1 2539.93
   148.6 2537.94   217.2 2537.56   249.3 2539.25   270.4 2537.99   291.4 2539.42
   308.3 2535.51   337.7 2534.85   354.5 2534.72   382.6 2535.08   413.5 2535.14
   436.4 2540.95   450.3 2540.81   464.1 2543.34   487.5 2540.36   505.7 2547.24
   535.9 2562.75   556.6 2569.24   566.6 2570.84   607.9  2573.4   670.1 2573.03
#Mann= 5 ,-1,0
       0      .1       0  297.66     .12       0  307.66      .1       0
   337.7    .045       0   382.6      .1       0
#XS Ineff= 2 , 0
                          466.14         2556.81
Permanent Ineff=
       F       F
Bank Sta=337.7,382.6
XS Rating Curve= 0 ,0
Exp/Cntr(USF)=0,0
Exp/Cntr=0.3,0.1

Type RM Length L Ch R = 1 ,62277   ,238.1,233.3,229.8
XS GIS Cut Line= 4
2356681.22553924700570.4611872952356822.84040825 700684.44388674
2356967.90929845700832.9667981382357140.61035822700957.311561169
#Sta/Elev= 30
       0 2615.14    55.4  2583.1    75.7 2566.98    87.3 2559.13   112.8 2539.22
   120.7 2536.37   126.4 2535.37   137.3 2537.43   157.4  2537.9   171.9 2534.01
   191.7 2533.88   206.6 2533.78   270.9    2534   290.7 2535.08   300.2 2534.31
   322.6 2540.16   398.3 2540.16   437.7 2538.65   449.9 2542.96   453.8 2543.27
   461.4 2542.29   467.1 2543.04     470 2544.29   478.8 2550.12   498.6 2558.97
   507.2 2561.76   518.7 2564.14   547.2 2567.97     582 2569.31   602.2 2571.87
#Mann= 3 ,-1,0
       0      .1       0   191.7    .045       0   270.9      .1       0
Bank Sta=191.7,270.9
XS Rating Curve= 0 ,0
Exp/Cntr(USF)=0,0
Exp/Cntr=0.3,0.1

Type RM Length L Ch R = 1 ,62043   ,178.8,174.5,170.2
XS GIS Cut Line= 3
2356487.71057459700798.4981837962356832.65811979  700898.1166559
2357095.82930729700996.248285137
#Sta/Elev= 30
       0 2625.21     9.7 2621.61    21.3 2615.18      38 2609.49    54.6 2601.39
    92.1 2587.79   117.1 2567.53   129.6 2554.83   137.9 2544.63   150.4 2533.53
   154.5 2532.56   170.5 2532.42   204.5 2532.42   212.5 2532.28   222.2 2532.57
   235.1 2536.16   275.3 2538.52   287.8 2537.09   362.8 2538.64   379.9 2537.46
   413.9 2539.05   452.4 2538.84     473 2537.34   490.9 2538.35   503.7 2542.74
   516.5 2543.31   533.6 2553.39   541.4  2555.6   576.2 2557.86   639.9 2566.46
#Mann= 3 ,-1,0
       0      .1       0   170.5    .045       0   204.5      .1       0
Bank Sta=170.5,204.5
XS Rating Curve= 0 ,0
Exp/Cntr(USF)=0,0
Exp/Cntr=0.3,0.1

Type RM Length L Ch R = 1 ,61869   ,307.2,297.2,282.3
XS GIS Cut Line= 2
2356460.16818274 701016.029921492357106.07014627701033.300027466
#Sta/Elev= 30
       0 2658.72      12 2647.68      24 2639.19    39.9 2625.42    56.4 2614.21
      68 2605.22   128.1 2566.12   140.1 2553.17   152.1 2541.63   156.1 2536.42
   160.1 2533.04   176.1 2531.51   220.1 2531.67   264.1 2536.77   280.1 2537.36
   304.1 2535.83   320.1 2537.27     336 2536.66   364.1 2533.42   384.1 2537.02
   480.2 2538.31   492.2 2541.94   504.2 2542.21   508.2 2543.33   520.2 2550.75
   528.2 2552.74   544.2 2554.64   599.1    2558   620.8 2560.62   646.1 2565.24
#Mann= 3 ,-1,0
       0      .1       0   176.1    .045       0   220.1      .1       0
Bank Sta=176.1,220.1
XS Rating Curve= 0 ,0
Exp/Cntr(USF)=0,0
Exp/Cntr=0.3,0.1

Type RM Length L Ch R = 1 ,61572   ,179.2,172.4,169.6
XS GIS Cut Line= 2
2356574.15088219 701413.242358952357068.07591312701102.380451372
#Sta/Elev= 30
       0  2713.1     2.4 2711.07    13.1  2694.9      45 2672.96    59.1 2664.87
    92.2 2639.58   111.1 2622.01   123.3 2614.19   153.6 2590.17   201.7 2547.48
   215.1  2530.9   230.7 2529.68     234 2529.59   265.5 2529.74   295.4 2534.75
     309 2534.53   323.8 2536.67   356.9 2535.03   375.8 2531.12   399.4 2537.84
   413.4 2538.16   441.9  2534.5   451.4  2534.9   462.7 2536.88   477.2 2542.18
   489.2 2542.01   498.7 2547.69   517.6 2552.57     527 2551.41   583.6 2554.66
#Mann= 3 ,-1,0
       0      .1       0   230.7    .045       0   265.5      .1       0
Bank Sta=230.7,265.5
XS Rating Curve= 0 ,0
Exp/Cntr(USF)=0,0
Exp/Cntr=0.3,0.1

Type RM Length L Ch R = 1 ,61399   ,347.1,339.4,330.5
XS GIS Cut Line= 3
2356817.29568534701504.1510215962357095.27549389 701194.12289319
2357139.50624665701120.612982426
#Sta/Elev= 30
       0  2627.8    10.3 2620.72    20.1  2611.3    25.5 2607.93    46.6  2589.5
      58 2581.11    73.8 2567.75    79.2  2562.8    84.6 2556.42    94.8    2542
   106.1 2531.37   111.4 2529.39   132.9 2528.93   154.3 2528.59   165.2  2528.7
   186.7 2529.62   196.8  2532.2     214 2535.07   229.6 2534.76     256  2538.2
   309.9  2535.3   332.7 2536.48   347.8 2540.91   352.6 2540.51   363.9 2538.03
   369.3 2540.17   375.8 2541.56   405.8  2544.8   452.7 2551.22   502.2 2563.45
#Mann= 3 ,-1,0
       0      .1       0   132.9    .045       0   165.2      .1       0
#XS Ineff= 2 , 0
                          347.99         2552.56
Permanent Ineff=
       F       F
Bank Sta=132.9,165.2
XS Rating Curve= 0 ,0
Exp/Cntr(USF)=0,0
Exp/Cntr=0.3,0.1

Type RM Length L Ch R = 1 ,61060   ,241.1,236.3,230.9
XS GIS Cut Line= 2
2357195.87469735701648.1158002312357323.62041701701153.592988872
#Sta/Elev= 30
       0 2609.74    19.1 2596.08      32 2588.66    48.5 2574.62    98.1 2535.32
   102.2 2530.65   106.3 2528.08   118.7 2527.29     160    2527   163.5 2527.03
   184.8 2527.33   188.9 2527.94   197.2 2531.64   213.7 2530.78     222 2532.88
     239 2534.64   250.9 2533.93   263.3 2535.04     284 2534.91   292.2 2536.53
   333.5 2539.65   354.2 2539.02   391.4 2540.51   416.2 2546.46   432.8 2552.02
   449.3 2559.05   461.6 2562.54   469.9 2563.76   478.1 2566.44   510.8 2570.34
#Mann= 3 ,-1,0
       0      .1       0   118.7    .045       0   163.5      .1       0
Bank Sta=118.7,163.5
XS Rating Curve= 0 ,0
Exp/Cntr(USF)=0,0
Exp/Cntr=0.3,0.1

Type RM Length L Ch R = 1 ,60824   ,356.3,352.3,348.6
XS GIS Cut Line= 2
2357461.83432938701699.9261181612357474.16922923701194.001760533
#Sta/Elev= 30
       0 2608.96    18.8 2596.94    30.8 2591.69    38.8  2587.3   102.8 2546.84
   114.8 2541.21   122.8 2535.32   134.8 2527.75   138.8 2526.38   150.8 2525.82
   154.8 2525.72   194.8 2525.92   222.8 2525.96   234.8 2530.61   246.8 2530.41
   266.7 2531.69   274.8 2532.97   282.3 2533.48   294.8 2532.69   313.5 2534.89
   338.8 2536.02   369.5 2535.27   382.9 2535.48   399.5  2537.2   422.9 2538.54
   458.9 2553.13   474.9  2561.5   478.9 2562.54   498.9 2570.47   506.1 2571.88
#Mann= 3 ,-1,0
       0      .1       0   150.8    .045       0   194.8      .1       0
#XS Ineff= 2 , 0
                          342.23         2546.26
Permanent Ineff=
       F       F
Bank Sta=150.8,194.8
XS Rating Curve= 0 ,0
Exp/Cntr(USF)=0,0
Exp/Cntr=0.3,0.1

Type RM Length L Ch R = 1 ,60471   ,239.8,240.6,240.7
XS GIS Cut Line= 2
 2357844.2377369  701673.65704932357767.21885161701171.991126036
#Sta/Elev= 30
       0 2581.89    12.6 2577.15    24.8 2575.14    32.9 2572.86    69.3 2559.05
   113.8 2544.56   138.1  2534.6   158.3 2524.25   170.5 2523.68   190.7 2523.54
   214.5 2523.72   231.2  2524.1   242.5 2528.14   256.6 2529.79   267.6 2529.01
   279.7    2530     300 2529.28   312.1  2531.6   337.3 2533.23   409.2  2532.8
   421.4 2533.52   437.5 2536.95   449.7 2537.79   453.7 2539.49   465.9  2548.1
     478 2555.04   486.1 2561.56   494.2 2570.33   498.2  2573.2   507.5 2577.33
#Mann= 3 ,-1,0
       0      .1       0   170.5    .045       0   214.5      .1       0
#XS Ineff= 2 , 0
                          352.06         2539.79
Permanent Ineff=
       F       F
Bank Sta=170.5,214.5
XS Rating Curve= 0 ,0
Exp/Cntr(USF)=0,0
Exp/Cntr=0.3,0.1

Type RM Length L Ch R = 1 ,60231   ,238.2,234.5,231
XS GIS Cut Line= 2
2358075.65715698701604.4840865122358004.46083004701132.818869952
#Sta/Elev= 30
       0 2558.84     7.4 2557.02    16.5 2556.29    48.1 2549.59    68.1 2547.07
    88.3 2541.87    96.4 2540.67   114.1 2534.41   124.7 2532.26   136.8 2524.53
   140.9 2523.34   144.9 2523.26   201.6 2522.96   202.8 2522.97   216.9 2523.28
   229.9 2526.24     242 2526.96   254.2 2528.86   286.5 2525.54   306.7 2527.54
   363.4 2530.87   379.6 2529.55   403.8 2530.37     416 2534.16   424.1 2535.58
   436.2 2543.39   444.3 2545.19   456.4 2554.57   464.5 2559.48     477 2568.57
#Mann= 3 ,-1,0
       0      .1       0   144.9    .045       0   202.8      .1       0
Bank Sta=144.9,202.8
XS Rating Curve= 0 ,0
Exp/Cntr(USF)=0,0
Exp/Cntr=0.3,0.1

Type RM Length L Ch R = 1 ,59996   ,195,183.7,178.1
XS GIS Cut Line= 2
2358329.29817828701558.4586667772358182.44950004701046.527857897
#Sta/Elev= 30
       0 2574.67    42.9 2560.35    47.1 2559.98    55.4 2557.43    67.9 2552.54
      97 2543.68   115.1 2539.09     122 2535.48   134.5 2523.84   155.3 2522.87
   209.4 2522.92   234.4 2522.65   251.1 2525.14     276 2526.05   300.9 2524.77
   317.6 2524.84   331.8 2526.27   367.5 2525.23   392.5 2532.02     405 2531.74
   409.1 2533.75   417.5  2541.3   434.1 2551.51   463.2 2571.75   475.7 2578.09
     484 2583.14   496.5 2588.93   504.9 2590.76   513.2 2594.55   532.6 2599.19
#Mann= 3 ,-1,0
       0      .1       0   155.3    .045       0   209.4      .1       0
Bank Sta=155.3,209.4
XS Rating Curve= 0 ,0
Exp/Cntr(USF)=0,0
Exp/Cntr=0.3,0.1

Type RM Length L Ch R = 1 ,59812   ,260.1,253.3,247.3
XS GIS Cut Line= 2
 2358561.8085855 701533.983887072358312.98165848  701054.6861178
#Sta/Elev= 30
       0 2615.76    13.7 2612.08    81.7 2583.83   109.1 2570.27   122.6 2562.02
   163.2  2545.3   172.2 2536.55   181.2 2523.94   185.7 2521.56   199.2 2522.57
   237.9 2521.24   262.9 2522.99   283.6 2521.57   307.4 2520.31   311.9  2521.4
   320.9 2524.06   329.9 2523.98   343.4 2526.23   360.8 2527.27   406.5 2523.69
     420 2529.41   433.6 2530.15   442.6 2536.67   458.7 2545.66   463.7 2549.81
   476.5 2564.37   497.3 2577.96   505.7 2580.85   528.2 2584.73     540 2584.97
#Mann= 3 ,-1,0
       0      .1       0   283.6    .045       0   311.9      .1       0
Bank Sta=283.6,311.9
XS Rating Curve= 0 ,0
Exp/Cntr(USF)=0,0
Exp/Cntr=0.3,0.1

Type RM Length L Ch R = 1 ,59559   ,223,222.5,222.7
XS GIS Cut Line= 2
2358755.56725819701295.3547849232358488.38424638701013.894818287
#Sta/Elev= 30
       0    2580     4.9 2576.18    16.5 2568.38      34 2557.56    51.4 2545.08
    74.7 2529.53    85.7 2521.25    91.6 2519.83   113.3 2519.91   150.2 2519.75
   165.2 2520.27     185 2523.15   190.5 2523.46     202 2523.58   212.6 2522.26
   218.1 2522.42   233.1  2524.4   243.1 2523.32   254.8 2522.95   267.7 2523.42
   272.7 2524.75   281.2 2529.01   295.4 2530.91   303.9  2535.5   322.9 2541.74
   340.6 2549.82   350.5 2552.54   359.3 2555.97   382.6 2560.78   388.1 2562.37
#Mann= 3 ,-1,0
       0      .1       0   113.3    .045       0   150.2      .1       0
Bank Sta=113.3,150.2
XS Rating Curve= 0 ,0
Exp/Cntr(USF)=0,0
Exp/Cntr=0.3,0.1

Type RM Length L Ch R = 1 ,59337   ,212.1,216.5,217.6
XS GIS Cut Line= 2
2358927.54113341701152.1483618122358663.92389305700879.164011389
#Sta/Elev= 30
       0 2595.48    16.4 2586.09    22.1 2582.22    26.4 2577.72    35.6 2561.59
    38.4 2557.66    45.2 2552.33    50.9 2547.04    62.4 2538.87    80.9 2528.47
    86.5 2524.67    92.2 2522.09     112  2520.5     120 2518.93   131.5 2518.72
   148.7 2519.59   189.1 2522.39   202.5  2521.3   225.1  2524.4   242.1 2522.66
   259.1 2522.67     271 2525.34   281.7 2529.34   292.8 2529.72   304.3 2533.94
   315.7 2534.84     327 2536.57   337.8 2539.69   348.9 2539.69   379.5 2543.79
#Mann= 3 ,-1,0
       0      .1       0     112    .045       0   148.7      .1       0
Bank Sta=112,148.7
XS Rating Curve= 0 ,0
Exp/Cntr(USF)=0,0
Exp/Cntr=0.3,0.1

Type RM Length L Ch R = 1 ,59120   ,207.5,198.1,191.3
XS GIS Cut Line= 2
2359078.75305301701019.6706623422358861.97136296700764.082373466
#Sta/Elev= 30
       0 2584.53      19 2574.82    22.5 2572.54    29.5  2566.3      40 2556.11
    45.2 2551.62    57.5 2542.37    80.2 2527.61    87.2 2524.37    96.7 2522.12
   105.8 2519.07   111.4 2518.35   118.7 2518.25   173.9 2518.19   181.6 2518.15
   199.4 2518.36   202.6 2518.75   213.1 2521.97   218.3 2522.07   226.6 2521.38
     242 2523.21   245.2 2523.16   256.2 2521.45   260.3 2521.42   284.6 2525.92
   291.7 2528.29   298.7 2529.69   312.9 2530.58     330 2530.71   335.1 2531.36
#Mann= 3 ,-1,0
       0      .1       0   118.7    .045       0   173.9      .1       0
Bank Sta=118.7,173.9
XS Rating Curve= 0 ,0
Exp/Cntr(USF)=0,0
Exp/Cntr=0.3,0.1

Type RM Length L Ch R = 1 ,58922   ,201.7,200.1,199.4
XS GIS Cut Line= 2
2359226.73589618700828.4856475022358896.88032605700632.083094294
#Sta/Elev= 30
       0 2583.05    16.9 2578.31    30.9 2572.03    35.6 2569.23    49.5 2556.45
    61.2  2546.4    72.8  2533.6    82.1 2525.16    86.8 2519.93    91.4 2517.72
   100.3 2517.31   105.4  2517.3   147.2 2517.34   161.8 2517.67   175.2 2520.08
   214.4 2520.02   225.4 2522.89   231.9 2523.27   255.2  2521.3   269.8 2521.32
   275.7 2522.36     287 2526.95   301.9 2530.53   328.9 2530.99   333.5 2531.94
   342.8 2530.37   351.5 2530.15   361.4 2532.61   370.8 2532.44   383.9 2533.65
#Mann= 3 ,-1,0
       0      .1       0   100.3    .045       0   147.2      .1       0
Bank Sta=100.3,147.2
XS Rating Curve= 0 ,0
Exp/Cntr(USF)=0,0
Exp/Cntr=0.3,0.1

Type RM Length L Ch R = 1 ,58722   ,263.1,253.6,253.1
XS GIS Cut Line= 2
2359319.90120988700642.1550200992358972.41976959700465.896318503
#Sta/Elev= 30
       0 2562.88      11 2557.79    15.4 2554.79    22.1    2549    31.1  2539.1
    44.5 2526.32    53.5 2520.65      58 2519.47    71.5 2519.45    83.8 2516.44
    92.8 2516.48   102.9 2516.24   161.2 2516.59   179.1 2516.75   183.6 2518.04
   187.8 2520.47     191 2521.53     206  2523.1     224 2522.77   244.5 2520.94
   273.3 2521.24   286.7  2525.8   300.2  2528.9   321.9 2530.21   331.6 2529.71
   345.1 2530.43   357.6 2531.56   366.5 2533.68   380.9 2534.47   389.6 2535.69
#Mann= 3 ,-1,0
       0      .1       0    92.8    .045       0   161.2      .1       0
Bank Sta=92.8,161.2
XS Rating Curve= 0 ,0
Exp/Cntr(USF)=0,0
Exp/Cntr=0.3,0.1

Type RM Length L Ch R = 1 ,58468   ,86.7,112.7,124.2
XS GIS Cut Line= 5
2359422.75204826700449.2364511712359411.08346215700376.468841737
2359234.42561123700347.0258665822359176.76645155700358.066982265
2359087.79611504700303.711915549
#Sta/Elev= 30
       0 2541.38    12.2 2540.98    36.5 2534.84    44.6 2530.97    52.7  2526.1
    61.7 2523.46    64.9 2522.81    73.7 2523.65    92.7 2523.39    96.9 2522.56
     105 2517.32   109.1  2516.2   125.3 2515.91   141.4 2515.82   166.7 2515.95
   186.1 2516.44   190.3 2517.59   198.3 2518.37   210.5 2522.64   222.6 2523.71
   283.6 2525.45   311.5 2525.55   318.4 2524.88   321.6 2525.45   335.6 2533.31
   338.8 2533.94   376.6  2536.7   397.6 2537.28   408.6 2536.61   415.8 2537.95
#Mann= 3 ,-1,0
       0      .1       0   125.3    .045       0   166.7      .1       0
Bank Sta=125.3,166.7
XS Rating Curve= 0 ,0
Exp/Cntr(USF)=0,0
Exp/Cntr=0.3,0.1

Type RM Length L Ch R = 1 ,58356   ,280.2,320.4,339.4
XS GIS Cut Line= 4
2359435.72835665700475.9682443082359460.90817116700372.731004802
2359382.85074617 700241.795969332359322.41919133700045.393416122
#Sta/Elev= 30
       0  2542.1    31.7 2537.33    39.9  2534.5    48.2 2533.87    60.5 2529.87
    72.9 2523.72    93.5 2524.12   105.8 2521.63   126.9 2521.54   147.7 2520.03
   166.3 2520.22   170.7 2519.47   176.5 2516.52   182.3 2515.65   231.9 2515.58
   234.8 2515.49   263.5 2518.96   277.3 2518.87   286.9 2521.14     297 2522.31
   326.3 2520.67   334.7 2523.38   368.2 2531.25   386.1 2538.48   397.5 2541.12
   405.8 2544.45   418.2 2546.78   426.7 2550.32     447 2554.44   464.2 2556.27
#Mann= 3 ,-1,0
       0      .1       0   182.3    .045       0   231.9      .1       0
Bank Sta=182.3,231.9
XS Rating Curve= 0 ,0
Exp/Cntr(USF)=0,0
Exp/Cntr=0.3,0.1

Type RM Length L Ch R = 1 ,58035   ,334,380.3,391.7
XS GIS Cut Line= 2
2359447.71587218700533.5802992242359844.99739007 700088.73690948
#Sta/Elev= 30
       0 2542.65    26.1 2536.22    36.7 2536.09    54.7 2530.35   105.4 2520.79
   133.8 2523.61   147.9 2522.71   218.7 2522.39   225.8  2523.2   294.9 2517.39
   311.6 2519.78     317 2519.57   326.4 2518.49   337.7 2514.88   351.9 2513.83
   365.2 2513.33   397.2 2513.41   408.1 2514.62   414.2 2518.77   424.2 2530.94
   434.9 2540.56   445.1 2551.65   472.5 2588.66   490.7 2605.25   499.3 2610.25
     519 2627.79   531.5 2634.76   541.1 2642.46   574.4 2663.86   596.4 2679.38
#Mann= 3 ,-1,0
       0      .1       0   351.9    .045       0   397.2      .1       0
Bank Sta=351.9,397.2
XS Rating Curve= 0 ,0
Exp/Cntr(USF)=0,0
Exp/Cntr=0.3,0.1

Type RM Length L Ch R = 1 ,57655   ,249.5,254,250
XS GIS Cut Line= 3
2359512.06428705700541.9735707282359671.53644564700550.366842233
2359878.57047609700651.086100288
#Sta/Elev= 30
       0 2527.45     9.4  2525.3    16.1 2524.53    36.2 2518.95    44.2 2517.81
    68.2 2518.18    76.2 2520.39    80.2 2520.89   104.3 2516.72   140.3  2515.3
   148.3 2513.78   160.4 2513.21   171.3 2511.03   211.8 2510.53   218.2 2510.78
   222.7 2511.64   230.1 2516.17     252 2540.37     258 2545.98   262.7 2549.91
   271.6  2555.4   280.5 2562.62   305.9 2581.12   319.6 2588.39   335.8 2599.18
   344.8 2603.98   360.6  2615.9   369.5 2619.41   377.7 2624.43   389.9 2629.74
#Mann= 4 ,-1,0
       0      .1       0   171.3    .045       0   211.8      .1       0
  299.69     .06       0
Bank Sta=171.3,211.8
XS Rating Curve= 0 ,0
Exp/Cntr(USF)=0,0
Exp/Cntr=0.3,0.1

Type RM Length L Ch R = 1 ,57401   ,216.4,212.9,212.9
XS GIS Cut Line= 2
2359355.38988563700653.8838574562359791.84000387700877.704430912
#Sta/Elev= 30
       0 2570.24     9.9 2568.55    41.3 2558.79    63.8 2553.34    89.2 2543.75
   101.1 2540.99   113.3 2534.67   122.3  2531.2   130.8 2526.42   135.7 2523.09
   144.7 2514.81   147.5 2513.36   169.4 2509.51   185.2 2509.21     211 2509.55
   252.6 2512.56   266.1 2514.44   284.1 2513.66   297.6 2517.82   311.1 2518.73
     320 2521.13   360.5    2544   374.5 2550.49   384.2 2557.48     401 2566.67
   436.7 2590.21   454.3 2600.31   472.9  2612.4   484.4 2620.89   490.5 2624.16
#Mann= 3 ,-1,0
       0      .1       0   169.4    .045       0     211      .1       0
Bank Sta=169.4,211
XS Rating Curve= 0 ,0
Exp/Cntr(USF)=0,0
Exp/Cntr=0.3,0.1

Type RM Length L Ch R = 1 ,57188   ,291.5,291.6,291.6
XS GIS Cut Line= 2
2359257.46838475 700849.726859232359696.71626015701053.963132509
#Sta/Elev= 30
       0 2585.04    16.2  2584.3      25 2582.15    42.7 2576.25    55.8 2570.83
    74.6 2558.58    86.8  2551.9    95.6 2545.57   104.4  2538.5   122.1 2514.95
   128.1 2510.29   130.9 2508.96   135.3 2508.36     153 2508.12   188.3 2508.41
   227.5 2509.65   241.2 2512.37     250 2512.15   260.6 2513.61   275.6 2513.72
   289.7  2514.9   307.4 2517.43   320.8 2517.83   349.7 2523.21   396.1 2542.13
   413.2 2551.63   432.2 2560.53   457.3 2575.95   470.6 2583.38   484.4 2590.09
#Mann= 3 ,-1,0
       0      .1       0   135.3    .045       0   188.3      .1       0
Bank Sta=135.3,188.3
XS Rating Curve= 0 ,0
Exp/Cntr(USF)=0,0
Exp/Cntr=0.3,0.1

Type RM Length L Ch R = 1 ,56896   ,273,274,272
XS GIS Cut Line= 2
2359078.41192598701087.5362185272359540.04185873701302.963520479
#Sta/Elev= 30
       0 2601.32      24 2596.31    37.3 2591.66    50.5 2588.92    59.7 2585.79
    81.4 2575.93    90.2 2570.82   101.9 2565.34     129 2549.46     135 2546.99
   138.8 2544.34   156.4 2529.03   178.5 2516.24   187.3 2510.12   196.2 2507.27
   230.9 2506.68   249.1 2507.26   276.4 2508.16   291.5 2507.76   306.5 2510.19
   319.8  2510.7   346.2 2516.26   360.7 2516.56   368.3 2518.33   408.9  2522.4
     439 2526.41   443.4 2527.44     461 2534.69   486.3 2542.23   509.4 2551.96
#Mann= 4 ,-1,0
       0      .1       0   196.2    .045       0   249.1      .1       0
     490     .06       0
Bank Sta=196.2,249.1
XS Rating Curve= 0 ,0
Exp/Cntr(USF)=0,0
Exp/Cntr=0.3,0.1

Type RM Length L Ch R = 1 ,56622   ,242,242.6,245.8
XS GIS Cut Line= 3
2358934.00871202701323.3869524832359228.11148064701456.478666125
     2359426.628      701582.618
#Sta/Elev= 30
       0 2604.84    15.5 2600.22    33.1 2590.97    50.7 2583.61    66.5 2574.35
    72.6 2569.32    84.6 2563.01   114.8  2542.1   125.3 2536.83   145.1 2524.62
   173.6 2513.29   186.8 2506.43   191.2  2505.3   204.3 2504.87   208.5  2504.9
     269 2505.18   296.5 2507.61   341.8 2508.89   356.1 2506.94   366.8 2510.32
   372.6 2510.42   381.3 2508.97   392.9 2512.44   408.2 2512.73   422.4 2516.03
   433.5 2519.87   450.9 2528.91   493.5 2554.39     503 2558.98     558 2592.03
#Mann= 5 ,-1,0
       0      .1       0   208.5    .045       0     269      .1       0
     300     .06       0  412.82      .1       0
Bank Sta=208.5,269
XS Rating Curve= 0 ,0
Exp/Cntr=0.3,0.1

Type RM Length L Ch R = 1 ,56380   ,92.5,100.2,103.9
XS GIS Cut Line= 2
 2358746.6569149 701482.218501222359324.69612729701785.452186405
#Sta/Elev= 30
       0    2608     6.2 2606.92    15.3 2602.18    28.8 2599.35    46.9 2591.71
      65  2586.2    74.4 2581.13    87.5 2577.19   110.1 2567.77   130.7 2562.12
   155.3 2552.77     184 2538.45   195.8 2533.84     205 2527.66   227.6 2518.51
   254.7 2504.24   268.2 2502.82   272.1 2502.79   326.3 2503.18     347 2504.86
   385.7 2505.14   403.3 2507.39   417.3 2506.74     430 2508.73   448.9 2505.06
   457.9 2505.91   471.5 2511.99   492.2 2525.36   557.4 2571.88   652.7 2626.74
#Mann= 4 ,-1,0
       0      .1       0   268.2    .045       0   326.3     .06       0
     520      .1       0
Bank Sta=268.2,326.3
XS Rating Curve= 0 ,0
Exp/Cntr(USF)=0,0
Exp/Cntr=0.3,0.1

Type RM Length L Ch R = 1 ,56280   ,403.6,398.7,401
XS GIS Cut Line= 2
2358764.57236074701545.7401858812359182.68585037701888.840511876
#Sta/Elev= 30
       0 2583.88      18 2576.58      42 2569.58    50.5 2564.88    61.6 2563.19
    71.9 2557.86    87.4  2554.1     103  2548.2   131.5 2531.77   149.5  2525.2
   165.1 2517.11   186.9 2512.63   201.3  2508.3   209.6 2503.57   216.8 2502.53
   242.7  2502.3   268.6 2502.55   280.7 2502.44   294.4 2504.95   314.8 2504.71
     329 2505.91   354.6 2506.46   366.9  2505.1   387.6 2510.43   391.5 2512.74
   402.9 2523.92   411.4 2529.95     437 2542.17   485.9 2571.27   540.9  2601.4
#Mann= 5 ,-1,0
       0      .1       0   216.8    .045       0   268.6      .1       0
     320     .06       0     440      .1       0
Bank Sta=216.8,268.6
XS Rating Curve= 0 ,0
Exp/Cntr=0.3,0.1

Type RM Length L Ch R = 1 ,55881   ,265.8,256.2,253.3
XS GIS Cut Line= 3
2358530.32407545701825.6878567242358685.49522354701967.245781736
2358920.16874541702186.435829788
#Sta/Elev= 30
       0 2545.47    28.9 2535.45    45.8 2531.74    60.4 2525.39    74.6 2522.55
   105.4 2512.17     117  2506.3   122.7 2504.91   175.8  2506.6   193.5 2505.36
   208.3  2501.8   224.7 2503.53   241.1 2501.53   255.8 2503.93     263 2502.11
   283.2 2500.72   323.2 2501.71   335.9 2500.57   359.4    2500   371.1 2500.64
   388.8 2506.85   399.8 2509.39   405.3 2512.11   425.6 2532.36     434 2542.24
   439.7 2546.88   445.4 2550.13   476.4 2566.47   513.3 2579.72   531.2 2587.76
#Mann= 5 ,-1,0
       0      .1       0   335.9    .045       0   371.1      .1       0
  380.04     .06       0  520.04      .1       0
Bank Sta=335.9,371.1
XS Rating Curve= 0 ,0
Exp/Cntr(USF)=0,0
Exp/Cntr=0.3,0.1

Type RM Length L Ch R = 1 ,55625   ,195.7,202.7,193.4
XS GIS Cut Line= 4
2358299.77557798702036.7481111452358482.09623152702182.117394935
 2358772.9678902702339.6145510782358887.40330056 702409.43863968
#Sta/Elev= 30
       0 2542.68    31.2 2529.45    39.2 2527.14    56.8  2519.8    87.5 2510.46
    97.7 2506.03   116.2 2501.56   133.5 2500.38   142.9 2501.48   199.8 2501.43
   240.1 2503.41   303.8 2504.42     322  2503.7   335.6 2499.47   353.8 2499.39
   362.9 2499.32   402.2 2499.51   425.8 2500.08   431.7  2501.3   440.2 2505.01
   449.4 2506.29   453.9 2507.76   461.2 2511.95     476  2523.3   508.5 2540.44
   535.8 2557.16   549.4 2566.39     613  2591.8   652.1 2601.93     698 2608.52
#Mann= 4 ,-1,0
       0      .1       0   353.8    .045       0   402.2     .06       0
  613.95      .1       0
Bank Sta=353.8,402.2
XS Rating Curve= 0 ,0
Exp/Cntr=0.3,0.1

Type RM Length L Ch R = 1 ,55422   ,299.6,284.1,283.7
XS GIS Cut Line= 3
2358138.98263291702196.1003370022358315.49651878702306.635082816
2358647.15836195702486.680083395
#Sta/Elev= 30
       0 2565.69    13.3 2557.42      22  2553.8    48.6 2538.55    67.5 2529.91
    88.7 2518.71     109 2511.13   114.8 2507.56   124.1 2505.71   138.3 2499.23
   147.7 2498.86   158.4 2500.85   199.6 2500.28   213.6  2501.5   245.4 2501.32
   272.8 2502.56     291 2502.21   318.3 2499.03   345.6 2500.15   369.9 2498.38
     398 2498.17   427.5 2498.55   440.7 2499.08   449.6 2503.31   473.5 2510.95
   502.7 2525.26   523.8 2537.51   532.2  2540.9   557.3 2554.62   585.6 2567.49
#Mann= 5 ,-1,0
       0      .1       0  358.27     .06       0   369.9    .045       0
   427.5     .06       0  558.27      .1       0
Bank Sta=369.9,427.5
XS Rating Curve= 0 ,0
Exp/Cntr(USF)=0,0
Exp/Cntr=0.3,0.1
