HEC-RAS study GLADYFK.prj: GLADYFK

--- GLADYFK.g01 (geometry) --- (continued)

Type RM Length L Ch R = 1 ,55138   ,240.8,240.8,237.8
XS GIS Cut Line= 3
2357928.89514837702458.4422119532358463.39212335702669.706423906
2358574.20762613702683.378593468
#Sta/Elev= 30
       0 2625.21    16.4 2616.74      57 2592.02      68 2584.18    80.9 2579.57
   112.5 2558.56   137.2 2545.06   171.1 2522.91   205.7 2508.27   214.3 2501.06
   231.5 2497.89   240.1 2499.65   288.2 2499.76   308.9  2497.6   331.4  2497.1
   369.1 2496.77   410.1 2497.11     430 2497.19   445.5 2499.64   459.4 2505.48
   472.3 2506.95     481 2512.99   494.8 2519.22   506.8 2521.49   562.4 2537.92
   573.3 2539.62   599.7 2547.95   619.9 2550.29     636  2555.5   686.4 2560.96
#Mann= 5 ,-1,0
       0      .1       0   331.4    .045       0   410.1      .1       0
     420     .06       0     530      .1       0
Bank Sta=331.4,410.1
XS Rating Curve= 0 ,0
Exp/Cntr=0.3,0.1

Type RM Length L Ch R = 1 ,54897   ,171.8,162.7,151.2
XS GIS Cut Line= 4
2357927.03812095 702732.718284372358205.61131307702817.214430144
2358311.33977221 702836.89979012 2358525.3185339702779.475870641
#Sta/Elev= 30
       0 2593.02     5.4 2589.02    13.7 2584.72    30.4 2579.31    55.5 2569.15
     114 2530.82   126.6 2520.93   139.1 2508.29   151.7 2497.84   172.6  2495.6
   205.6 2495.74   218.5  2495.3   270.7 2495.46   293.3 2497.89   300.1 2500.28
   305.9 2500.98   342.5 2500.48     371 2503.45   399.5 2502.73   469.9 2506.12
   497.1 2514.04   527.9 2526.91   540.3 2528.88   548.6 2532.24     561 2534.95
   569.3 2538.37   577.6 2539.13   602.5 2545.23   611.3 2545.16   620.2  2547.3
#Mann= 5 ,-1,0
       0      .1       0   205.6    .045       0   270.7      .1       0
  311.11     .06       0  408.65      .1       0
Bank Sta=205.6,270.7
XS Rating Curve= 0 ,0
Exp/Cntr(USF)=0,0
Exp/Cntr=0.3,0.1

Type RM Length L Ch R = 1 ,54734   ,277.6,257.9,235.5
XS GIS Cut Line= 3
2357882.93181325702964.895023442 2358369.2624576702928.835743953
2358538.68883527702829.475639687
#Sta/Elev= 30
       0 2635.55    17.3 2623.66    29.3 2611.89    41.4 2603.16    65.4 2590.14
    81.5 2576.04    97.5  2564.5   109.5 2553.25   129.6 2541.46   141.6 2530.63
   157.6 2512.66   173.7 2498.47183.99712494.453242.39622494.351   249.9 2494.19
     278 2497.53   306.1 2495.01   322.1  2499.5   358.2 2498.73   398.3    2503
   462.5  2501.8   532.8  2504.3   542.1 2507.48   552.9 2508.56   569.9 2516.13
   583.1 2518.73   612.3 2530.26   626.9  2532.2   660.9 2540.76   684.1 2543.45
#Mann= 5 ,-1,0
       0      .1       0183.9971    .045       0242.3962      .1       0
     340     .06       0     440      .1       0
Bank Sta=183.9971,242.3962
XS Rating Curve= 0 ,0
Exp/Cntr(USF)=0,0
Exp/Cntr=0.3,0.1

Type RM Length L Ch R = 1 ,54476   ,149.2,148.9,149.4
XS GIS Cut Line= 3
2358088.80579049703316.7558492112358358.57080221703029.791808146
2358575.37415811702842.450804325
#Sta/Elev= 30
       0 2654.36    19.1 2641.05    48.8 2617.22      70 2604.73    81.3 2592.14
    95.5 2582.14   115.9 2565.52   131.2 2555.77   139.2 2548.11   150.9 2540.02
   191.7 2498.24   197.3 2495.09   211.5 2492.55     219  2492.3   261.9 2492.38
   268.1 2492.96   285.2 2496.78   327.5 2498.59   361.5 2502.66   384.5 2500.95
   411.8 2500.91   446.5 2503.19   496.4    2503   504.9 2505.64   514.5 2506.64
   547.7 2518.28   612.7 2533.77   623.3 2534.88   639.3  2540.1   680.4 2545.29
#Mann= 5 ,-1,0
       0      .1       0   211.5    .045       0   261.9      .1       0
     350     .06       0  493.85      .1       0
#XS Ineff= 2 , 0
                          365.23         2526.58
Permanent Ineff=
       F       F
Bank Sta=211.5,261.9
XS Rating Curve= 0 ,0
Exp/Cntr=0.3,0.1

Type RM Length L Ch R = 1 ,54328   ,219.4,209.1,198.7
XS GIS Cut Line= 2
2358202.46223007703425.7678944232358694.86749167702849.429917773
#Sta/Elev= 30
       0 2668.77    33.4 2641.35    44.2 2635.54    64.2 2620.04    95.3 2600.58
   115.1 2584.67   179.7 2538.54   190.2 2527.42   203.1 2516.43   211.6 2511.72
   232.3 2494.49   242.7 2492.63   292.1 2491.91   305.9 2491.98   332.2 2496.46
   390.3    2502   400.6 2500.69   416.4 2502.51   469.8 2501.04   505.8 2502.11
   560.5 2514.89   593.8 2520.13   600.5 2519.41   642.6 2528.47     657 2533.31
   668.4 2533.78   693.9 2540.84   732.1 2547.14   742.6 2551.41     758 2554.53
#Mann= 5 ,-1,0
       0      .1       0   242.7    .045       0   305.9      .1       0
     350     .06       0     480      .1       0
Bank Sta=242.7,305.9
XS Rating Curve= 0 ,0
Exp/Cntr(USF)=0,0
Exp/Cntr=0.3,0.1

Type RM Length L Ch R = 1 ,54118   ,313.3,306.6,298.6
XS GIS Cut Line= 3
2358457.25619076703592.264448922 2358632.7804663703146.064088602
2358768.95236796702882.244741836
#Sta/Elev= 30
       0 2707.37    46.3 2670.29    97.9 2634.27     128 2615.01   158.1 2592.43
   166.7 2584.97   180.5 2569.44   193.7 2546.94   213.9 2528.35     244 2506.31
   269.8 2491.78   285.4 2490.96   313.1 2490.73     347 2490.88   360.1 2491.77
     373  2494.8   398.8 2494.74   424.2 2500.23   534.5 2499.44     566 2501.85
   610.3 2513.58     643 2517.93     674 2526.41     683 2527.22   713.6 2537.93
   722.4 2543.01   732.1 2543.53   759.6 2555.57   768.6 2556.33   776.4 2559.48
#Mann= 5 ,-1,0
       0      .1       0   285.4    .045       0     347      .1       0
     360     .06       0     470      .1       0
Bank Sta=285.4,347
XS Rating Curve= 0 ,0
Exp/Cntr=0.3,0.1

Type RM Length L Ch R = 1 ,53812   ,178.3,173.2,166.2
XS GIS Cut Line= 2
2358845.94637875703543.2736954872358935.47460813702888.598518128
#Sta/Elev= 30
       0 2646.02    14.2 2634.01    22.3 2622.63    26.3 2618.98    46.5 2603.35
   127.3 2532.86   147.5 2511.84   159.6 2492.49   163.6 2489.53   183.8  2488.9
   232.2 2488.69   240.3 2488.57   256.5 2491.52   268.6 2490.69   292.8 2494.24
     313 2493.21   329.1    2498   361.4 2499.52   393.7 2499.77   405.8 2497.71
   470.4 2495.64   486.6 2497.41     527 2509.81   571.4 2528.95   583.5 2535.61
   595.6 2539.73   615.8 2550.61   631.9 2554.93   648.1 2563.12   660.8 2564.47
#Mann= 7 ,-1,0
       0      .1       0   183.8    .045       0   232.2      .1       0
     290     .06       0     390      .1       0     450     .06       0
     490      .1       0
#XS Ineff= 2 , 0
                          443.98         2520.03
Permanent Ineff=
       F       F
Bank Sta=183.8,232.2
XS Rating Curve= 0 ,0
Exp/Cntr(USF)=0,0
Exp/Cntr=0.3,0.1

Type RM Length L Ch R = 1 ,53639   ,306.4,304.2,304.6
XS GIS Cut Line= 3
2359069.61014073703534.2514739382359035.13291522703236.914470117
2359001.50030228 703008.32506852
#Sta/Elev= 30
       0 2611.83     9.1 2606.85    45.4 2590.13    53.4 2584.03    63.4 2579.19
    77.6 2570.48    85.6 2566.83   109.8 2549.52   121.9  2537.6   125.9  2534.9
     146 2517.76   174.2 2489.52   179.1 2487.99   226.6 2487.24   227.3 2487.26
   242.7 2487.54   258.8 2489.42   286.5 2490.63   299.1 2490.16   311.2 2493.35
   327.4 2492.59   339.5 2496.22   347.6 2495.97     384 2498.46   416.3 2497.09
   424.4 2497.55   448.7 2495.97   497.2 2496.35   517.4 2499.45   530.4 2505.33
#Mann= 5 ,-1,0
       0      .1       0   179.1    .045       0   227.3      .1       0
     280     .06       0  479.33      .1       0
Bank Sta=179.1,227.3
XS Rating Curve= 0 ,0
Exp/Cntr=0.3,0.1

Type RM Length L Ch R = 1 ,53334   ,195.2,190.3,187
XS GIS Cut Line= 2
2359366.32921204703406.1835942452359285.19425416702944.553661492
#Sta/Elev= 30
       0 2537.29    17.3 2530.71    33.5 2523.29    45.7 2519.19    74.1 2507.77
   104.9 2496.43   114.7  2492.4   122.9 2487.36   127.1 2486.13   140.9  2485.4
   187.8 2485.23     196 2485.34   216.3 2485.84   244.7 2490.14   273.1 2489.37
   285.3 2489.69   296.3 2492.79   301.6 2493.45   313.7 2492.66   338.1  2494.8
   350.3 2494.98   366.5 2493.95   374.7 2494.16   382.8 2493.22     399 2493.19
   431.5 2494.18   439.6 2495.17   451.8 2495.16   459.9 2499.96   468.7 2504.06
#Mann= 5 ,-1,0
       0      .1       0   140.9    .045       0     196      .1       0
     250     .06       0     350      .1       0
#XS Ineff= 2 , 0
                          370.83         2500.65
Permanent Ineff=
       F       F
Bank Sta=140.9,196
XS Rating Curve= 0 ,0
Exp/Cntr(USF)=0,0
Exp/Cntr=0.3,0.1

Type RM Length L Ch R = 1 ,53144   ,268.7,271.1,272.3
XS GIS Cut Line= 3
2359578.41079014703349.2413293922359459.92266088703024.780236969
2359390.69316956702826.393063586
#Sta/Elev= 30
       0 2539.12    29.8  2526.7    63.9 2510.85    89.5 2501.74   107.8  2497.8
   127.8 2492.32   149.1  2491.4   166.1 2486.25   178.9  2484.6   242.8 2484.29
   260.7  2485.3   272.6  2488.6   304.4 2488.82   323.7 2491.69   336.5 2490.78
   353.5 2492.06   374.7 2490.76   395.8 2490.84   412.8 2493.05     434  2494.5
   450.9 2497.52   467.9 2505.32   492.5 2519.51   498.8 2522.07     506 2527.13
   514.5 2531.49   522.9 2537.54   536.5 2544.29   544.1 2549.94   555.5 2554.98
#Mann= 4 ,-1,0
       0      .1       0   178.9    .045       0   242.8     .06       0
     310      .1       0
Bank Sta=178.9,242.8
XS Rating Curve= 0 ,0
Exp/Cntr=0.3,0.1

Type RM Length L Ch R = 1 ,52873   ,248.1,246.4,255
XS GIS Cut Line= 2
2359827.95914479703283.0822788442359640.50941452702661.980187504
#Sta/Elev= 30
       0 2551.22    14.5  2545.8    39.6 2532.61     119 2501.71   155.4 2491.06
     190 2484.41   198.4 2483.88   219.3 2483.27   258.1 2483.68   294.5 2483.68
   323.7  2487.5     353 2489.62   382.2  2488.9   418.6 2493.02     440 2500.08
   453.2 2506.55   465.8 2515.74   478.3 2519.18   486.7 2527.84     495 2533.16
   507.6 2544.21   515.9 2548.48   549.3 2575.27   565.7 2583.23   574.4 2590.43
   582.8 2593.94   599.5 2608.48     612  2612.6   641.3 2636.53   648.8 2640.27
#Mann= 5 ,-1,0
       0      .1       0   198.4    .045       0   258.1      .1       0
     340     .06       0     440      .1       0
Bank Sta=198.4,258.1
XS Rating Curve= 0 ,0
Exp/Cntr(USF)=0,0
Exp/Cntr=0.3,0.1

Type RM Length L Ch R = 1 ,52627   ,275.4,289.7,306.6
XS GIS Cut Line= 4
2359952.48361293703294.1560962442360027.95804888703148.770609943
2360002.33010598703035.4553391252359943.88616956702734.649254344
#Sta/Elev= 30
       0 2565.72    39.1 2559.04    65.8 2551.87   103.5 2536.44     137 2525.76
   160.7 2514.22   196.2 2494.48   224.9 2485.32   237.2 2484.27   278.2 2487.45
   290.5 2485.21   302.7 2485.54   333.2 2481.84   343.4 2481.58   396.1 2482.06
   412.7 2482.57   424.9 2484.68   433.1 2483.48   445.3 2488.65   457.5 2490.17
   473.8 2495.27   488.5 2505.32   502.7 2518.11   510.5 2526.71   526.8 2539.94
     539 2543.45     543 2546.06   551.2 2554.94   575.7 2575.53   586.4 2582.43
#Mann= 4 ,-1,0
       0      .1       0   333.2    .045       0   396.1     .06       0
  459.99      .1       0
Bank Sta=333.2,396.1
XS Rating Curve= 0 ,0
Exp/Cntr=0.3,0.1

Type RM Length L Ch R = 1 ,52337   ,184,187.2,191.5
XS GIS Cut Line= 2
2360096.32305959703290.2996139832360345.60322328702839.580934186
#Sta/Elev= 30
       0 2549.87    47.8 2541.36    65.5 2536.82    90.6 2528.74   100.8 2524.53
     111 2518.38   120.1 2514.32   133.8 2503.65   165.8 2488.28   188.7 2486.63
   203.8 2483.48   216.1 2482.09   248.1 2483.92   312.1 2484.48   321.3 2483.25
   330.5 2480.29   344.1 2479.06   346.8 2479.03   377.4 2479.38   385.2  2479.5
     399 2481.91   408.1 2486.08   421.2 2488.59   424.5 2490.33   454.3 2517.06
   462.8 2525.71   476.7 2536.37   487.3 2546.07   508.7 2560.78   515.1 2563.97
#Mann= 5 ,-1,0
       0      .1       0   344.1    .045       0   377.4      .1       0
     380     .06       0     490      .1       0
Bank Sta=344.1,377.4
XS Rating Curve= 0 ,0
Exp/Cntr(USF)=0,0
Exp/Cntr=0.3,0.1

Type RM Length L Ch R = 1 ,52150   ,316.8,327.4,346.2
XS GIS Cut Line= 3
2360105.81860293703379.1527815882360231.51159111703322.692361493
     2360585.147      702870.695
#Sta/Elev= 30
       0 2555.58    50.8  2545.6    85.9  2536.2   195.6 2514.49   215.9  2506.7
   236.2 2495.15   256.5 2486.33   301.8 2485.97   327.4 2483.42   342.9 2479.69
   359.6 2482.18   427.1 2482.85   449.5 2478.63   454.6  2478.6   495.2 2478.81
   508.9 2479.29   520.6 2486.06   535.9 2488.67   551.1  2505.4   561.3 2512.76
   571.4 2523.39   578.2 2528.65   586.6 2539.02   599.8 2552.18   625.7 2570.07
   658.2 2589.27   669.3 2598.44   686.4 2607.77   700.7 2619.15   711.7 2622.66
#Mann= 4 ,-1,0
       0      .1       0   449.5    .045       0   495.2     .06       0
  597.79      .1       0
Bank Sta=449.5,495.2
XS Rating Curve= 0 ,0
Exp/Cntr=0.3,0.1

Type RM Length L Ch R = 1 ,51822   ,241,246.4,263.9
XS GIS Cut Line= 2
2360229.77607652703423.752630907 2360831.5736434703285.263651081
#Sta/Elev= 30
       0 2529.49    96.9 2505.31   117.6 2502.36   154.2 2499.31   204.3 2485.77
     221 2482.88   236.4 2482.45   256.9 2477.41   281.6  2479.8   289.8  2481.7
   306.2 2482.64   326.7 2482.26   347.2 2476.89   363.7 2476.75   380.1  2476.5
   404.6 2476.76   421.7 2477.71   425.2 2478.88   433.4 2485.36   441.6 2486.19
   449.9 2490.56   464.6 2504.53   474.5 2512.72   491.3 2530.84   515.5 2554.57
   519.6 2557.77   531.9  2564.4   551.4 2581.44   589.4 2608.71   617.5 2626.75
#Mann= 5 ,-1,0
       0      .1       0   363.7    .045       0   404.6      .1       0
     470     .06       0     570      .1       0
Bank Sta=363.7,404.6
XS Rating Curve= 0 ,0
Exp/Cntr(USF)=0,0
Exp/Cntr=0.3,0.1

Type RM Length L Ch R = 1 ,51576   ,262.3,266.4,278.1
XS GIS Cut Line= 4
2360225.07066837703462.8869988042360362.39122219703498.004115016
2360481.13570485703547.7578330622360810.45790726703679.114666125
#Sta/Elev= 30
       0 2529.29    23.8 2523.94    44.5 2515.08    77.5 2504.87   131.2 2493.94
   148.6 2489.25   178.4 2486.42   191.4 2481.84   200.1 2481.62   209.7 2479.28
   234.7 2481.66   260.8 2481.97   273.8    2478   286.7 2475.98   295.9    2476
   308.2 2478.23   329.7 2474.59   338.4 2474.75   372.8 2474.98   394.3 2475.41
   398.6 2477.09   406.3 2482.96   415.9 2485.33   421.7 2489.42   450.3 2512.65
   498.7 2549.64   536.5 2581.55   584.9 2624.42   596.7 2638.08     625 2665.63
#Mann= 5 ,-1,0
       0      .1       0   338.4    .045       0   372.8      .1       0
  380.49     .06       0  490.49      .1       0
Bank Sta=338.4,372.8
XS Rating Curve= 0 ,0
Exp/Cntr=0.3,0.1

Type RM Length L Ch R = 1 ,51310   ,228.5,236.7,255.6
XS GIS Cut Line= 3
2360101.43260131703597.1724309662360305.38909887703697.891689021
2360572.29513272 703972.35166722
#Sta/Elev= 30
       0 2540.68      23 2532.77    34.9 2526.81    72.3 2514.03   123.5 2493.17
   145.8 2486.84   163.7 2484.86   232.1 2484.98   242.9 2483.47   262.9 2477.86
   291.2 2478.06   304.6 2473.36   310.2 2472.96   319.5 2472.98   373.2 2473.17
   399.4 2473.65   403.6 2475.54   410.6 2481.14   421.8 2482.75   427.3 2485.34
   443.9 2501.13   466.7 2520.32   488.7 2542.78   535.6 2586.14   564.2 2614.45
   583.6  2629.9   587.2 2636.19     591 2646.66   594.7 2654.65   610.3 2669.67
#Mann= 5 ,-1,0
       0      .1       0  307.47     .06       0   319.5    .045       0
   373.2     .06       0  447.47      .1       0
Bank Sta=319.5,373.2
XS Rating Curve= 0 ,0
Exp/Cntr(USF)=0,0
Exp/Cntr=0.3,0.1

Type RM Length L Ch R = 1 ,51073   ,167.8,165.4,160.7
XS GIS Cut Line= 2
2360117.38768709703674.5607180872360202.12111711 704012.46526155
#Sta/Elev= 30
       0 2508.79    15.1 2501.06    39.8 2491.93    48.1 2489.34    56.3 2485.62
    64.6 2484.34    76.9 2480.88    85.2 2479.33    89.3 2478.15    97.5 2477.77
   106.7  2476.5     114 2474.76   122.3 2471.84   131.9 2471.61   192.4 2471.44
   197.9 2471.43   208.9 2471.91   217.1 2473.52   229.5 2477.88   237.8 2478.41
   241.9 2479.16     246 2481.21   251.7 2485.42   261.6 2491.26   280.5 2499.75
   307.9  2514.5   323.9 2524.23   328.5 2526.46   336.7 2531.36   348.4 2537.58
#Mann= 3 ,-1,0
       0      .1       0   131.9    .045       0   192.4      .1       0
Bank Sta=131.9,192.4
XS Rating Curve= 0 ,0
Exp/Cntr(USF)=0,0
Exp/Cntr=0.3,0.1

Type RM Length L Ch R = 1 ,50908   ,137.8,128.4,123.3
XS GIS Cut Line= 2
2359884.88619649703612.2803196742360101.43260131704105.804684143
#Sta/Elev= 30
       0 2567.09    40.3 2563.42    62.1 2560.47      70 2557.87    75.2 2554.01
    88.2 2546.74    97.1 2540.75   103.4 2532.51   109.4 2526.62   118.9 2518.65
   130.7 2511.02   142.8 2500.94   149.5 2496.51   162.6 2490.98   176.2 2481.27
   184.4 2476.68   206.6 2470.44   219.4 2471.08     260 2470.49   267.3 2470.31
   302.4 2470.64   346.7 2473.24   359.2 2476.01   373.6 2476.95   385.4 2482.36
     416 2492.42   455.5 2508.67     486 2520.05   525.4 2536.64   538.9 2544.42
#Mann= 5 ,-1,0
       0      .1       0     260    .045       0   302.4      .1       0
     370     .06       0     480      .1       0
Bank Sta=260,302.4
XS Rating Curve= 0 ,0
Exp/Cntr(USF)=0,0
Exp/Cntr=0.3,0.1

Type RM Length L Ch R = 1 ,50779   ,216.2,212.2,205.5
XS GIS Cut Line= 2
 2359748.3817624703674.7564227912359976.34930994704076.664265134
#Sta/Elev= 30
       0  2564.7    22.2 2559.77    53.4 2550.84    80.9  2536.8    94.8 2526.92
   108.6 2513.71   113.2 2511.07   117.8  2507.2   127.8 2496.88   140.7 2484.62
   149.9 2477.22   153.6 2475.34   161.7 2473.24   168.3 2472.76   180.6 2473.41
   186.7 2472.02     210 2469.49   241.9 2469.44   280.4 2469.64   318.5 2471.44
   330.3 2471.04   347.7 2472.51   359.6 2475.47   375.3 2475.71   384.5 2479.14
   412.1 2485.84     430 2492.45   447.6 2500.01   456.4 2502.05   462.1 2504.26
#Mann= 5 ,-1,0
       0      .1       0     210    .045       0   280.4      .1       0
     320     .06       0     430      .1       0
Bank Sta=210,280.4
XS Rating Curve= 0 ,0
Exp/Cntr(USF)=0,0
Exp/Cntr=0.3,0.1

Type RM Length L Ch R = 1 ,50567   ,173.6,167.4,162.6
XS GIS Cut Line= 3
2359541.03345243 703714.473157382359605.11971327703888.004642673
2359842.86592564704188.305638533
#Sta/Elev= 30
       0 2568.19    48.1 2559.43    62.6 2555.99    79.3 2553.81     101 2546.71
   109.5 2542.24   130.8 2525.97   147.9 2514.91   159.2 2502.69   173.4 2491.65
   177.7 2487.05   186.5 2480.18   191.6 2477.22   196.7 2472.65   201.8 2470.25
   222.2 2471.91   298.7 2471.99   308.9  2469.1   324.7  2468.7   375.3 2468.34
   395.9 2468.56   415.8 2468.53     430 2469.75   434.8 2471.31   441.6 2475.81
   456.9 2477.61   497.7 2487.41   512.1 2489.74   538.5 2497.33     568 2507.12
#Mann= 4 ,-1,0
       0      .1       0   324.7    .045       0   395.9     .06       0
  514.99      .1       0
Bank Sta=324.7,395.9
XS Rating Curve= 0 ,0
Exp/Cntr=0.3,0.1

Type RM Length L Ch R = 1 ,50399   ,269,272.9,279.4
XS GIS Cut Line= 2
2359228.28189777703809.0049507422359731.87818805704269.080573957
#Sta/Elev= 30
       0 2563.21    53.6 2556.27   112.9 2550.57   135.3 2549.79   151.6 2548.13
   169.9 2543.12   175.6 2540.06     196 2525.58   201.9 2518.26   215.2 2498.83
   219.7 2493.96   227.4 2488.01   237.5 2477.52   243.5 2473.34   254.5 2469.56
   291.7 2469.67   314.6 2468.11   427.3 2470.55   453.1 2467.59   464.4 2467.15
     470 2467.04   526.7 2467.37   549.3 2468.28   552.2  2469.1   557.8 2474.53
   566.3 2477.33   586.1 2478.52   628.3 2490.49     650 2494.67   682.1 2504.58
#Mann= 4 ,-1,0
       0      .1       0   464.4    .045       0   526.7     .06       0
     650      .1       0
Bank Sta=464.4,526.7
XS Rating Curve= 0 ,0
Exp/Cntr(USF)=0,0
Exp/Cntr=0.3,0.1

Type RM Length L Ch R = 1 ,50127   ,297.2,289.9,283.6
XS GIS Cut Line= 4
2359210.97223409703934.1527214782359232.46259888  704099.8893768
2359310.51586743704216.0975171822359504.74136824704423.117685745
#Sta/Elev= 30
       0 2542.09    99.9 2527.01   128.7 2519.54   135.9 2515.98   152.3 2503.49
   164.3 2489.49   173.5 2479.99     181 2469.46   183.1 2467.63     188  2465.9
   205.3 2465.43   216.9 2466.35   260.2 2466.69   295.7 2464.93   319.6 2466.06
   344.6 2465.14   388.3 2465.31   399.6 2465.54   412.8 2471.39   418.3 2472.79
   426.5 2471.86   451.2 2472.64   462.2 2474.11   473.1 2476.96   490.2 2477.51
     506 2482.08   518.5 2484.18   529.8 2487.73     539 2489.24     591 2508.33
#Mann= 4 ,-1,0
       0      .1       0   344.6    .045       0   388.3      .1       0
  487.11     .06       0
Bank Sta=344.6,388.3
XS Rating Curve= 0 ,0
Exp/Cntr=0.3,0.1

Type RM Length L Ch R = 1 ,49837   ,176.8,178.9,182.7
XS GIS Cut Line= 2
2358877.00794221704222.4512878212359315.32323189704520.878719095
#Sta/Elev= 30
       0 2498.42      10 2496.37    41.7 2493.72    54.6  2491.1    95.8  2489.2
     120 2490.46     149  2488.3   175.4 2482.57   182.9 2478.72   197.4 2467.84
   211.9 2465.93   221.6 2463.61   236.1 2463.23   283.5 2463.01   286.4 2463.12
   313.5 2465.34   338.2 2465.23   364.1 2469.22   410.2 2469.31   421.7 2471.15
   431.3 2471.46   444.7 2476.58   453.4 2473.85   459.7 2473.41   464.9 2474.56
   473.2 2479.04     485 2480.79   502.3 2485.56   511.9 2486.76   530.3 2492.42
#Mann= 4 ,-1,0
       0      .1       0   236.1    .045       0   286.4      .1       0
     390     .06       0
Bank Sta=236.1,286.4
XS Rating Curve= 0 ,0
Exp/Cntr(USF)=0,0
Exp/Cntr=0.3,0.1

Type RM Length L Ch R = 1 ,49658   ,189.4,206.3,221.6
XS GIS Cut Line= 3
2358701.38909538 704294.052095972359063.78161967704571.109428909
2359224.86036931704640.866212686
#Sta/Elev= 30
       0 2513.25    13.6 2508.51    28.7 2506.96    58.9  2499.7    98.4 2492.63
   126.5 2490.29     144 2486.39   186.8 2479.99   246.8 2474.76   260.3 2471.29
   270.4 2465.98   275.3 2465.12   289.6 2463.45   300.6 2465.56   314.7  2466.2
   329.5 2463.14     341 2462.75   386.2 2462.64   416.4  2463.4   426.5 2462.73
   455.1 2464.01   485.4 2468.28   503.7 2464.46     522 2464.54   535.1 2469.16
   548.1 2470.52   574.3 2478.56   587.4 2481.04   604.8 2487.02   631.7 2499.61
#Mann= 4 ,-1,0
       0      .1       0     341    .045       0   416.4     .06       0
  616.17      .1       0
Bank Sta=341,416.4
XS Rating Curve= 0 ,0
Exp/Cntr=0.3,0.1

Type RM Length L Ch R = 1 ,49451   ,322.5,303.2,280.8
XS GIS Cut Line= 4
2358544.87277021704426.955401728 2358815.3226298704588.603593668
2358861.95191594704691.1880231692359160.37934721704772.012119139
#Sta/Elev= 30
       0 2513.83    27.1 2506.53    92.4 2493.53   143.6 2487.32   196.5 2478.85
   254.9 2474.99   272.4 2465.29   277.2 2463.96   295.7 2463.83   315.7 2461.37
   346.1 2461.51   394.8 2461.28   416.8 2461.63   438.4 2466.17   450.8 2466.34
   463.2 2468.66   467.4  2466.8   483.9 2465.76   493.2 2462.62   504.7 2464.61
   525.4 2464.83   562.7 2460.19     619 2467.78     629  2472.4   639.9 2474.95
     658 2482.84   670.4 2486.29     679 2490.99   720.2 2507.62   736.9 2516.24
#Mann= 5 ,-1,0
       0      .1       0   346.1    .045       0   394.8      .1       0
  477.76     .06       0  577.76      .1       0
Bank Sta=346.1,394.8
XS Rating Curve= 0 ,0
Exp/Cntr(USF)=0,0
Exp/Cntr=0.3,0.1

Type RM Length L Ch R = 1 ,49148   ,281.8,274.7,267.4
XS GIS Cut Line= 3
2358294.95280983704810.3911901672358818.37766824704836.465238152
2359129.55771091704864.275905212
#Sta/Elev= 30
       0 2551.46    21.2 2539.75    41.3 2532.67    57.3 2524.19    89.3 2510.74
   133.4 2496.26   185.5 2485.51   209.5 2484.36   257.5 2478.77   293.6 2477.34
   305.6 2474.65   317.6 2461.12   321.6 2459.05   331.9 2458.62   361.7 2458.38
   365.7 2458.48   397.7 2462.34   530.1 2462.39   578.1  2464.5   586.1 2460.52
   610.2 2463.58   622.2 2462.16   646.4 2463.37   670.5 2459.38   694.5 2459.51
   714.4 2469.99   734.7 2486.22   794.9 2517.79     807 2522.65   836.5 2527.86
#Mann= 5 ,-1,0
       0      .1       0   331.9    .045       0   365.7      .1       0
  614.07     .06       0  714.07      .1       0
Bank Sta=331.9,365.7
XS Rating Curve= 0 ,0
Exp/Cntr=0.3,0.1

Type RM Length L Ch R = 1 ,48874   ,235.7,230.1,222
XS GIS Cut Line= 2
2358408.09353087705210.3274088232359101.31558477704942.986168307
#Sta/Elev= 30
       0 2558.25    30.1 2542.48    81.4 2518.83    94.4  2511.7   146.4 2466.71
   154.4 2461.09   158.6 2459.68   274.5 2460.39   291.6 2457.77   325.6 2457.37
   381.2 2457.12   390.2 2457.17   415.9    2461     446 2461.69   467.4 2460.36
   484.5 2460.99     496 2456.28     506 2455.68   517.6 2457.87   526.9 2456.61
   531.7 2458.89   540.3 2465.21   557.9  2464.8   570.3 2468.16   578.9 2473.69
   604.6 2496.92   625.9 2505.31   650.7 2513.18     686 2520.85     743  2527.1
#Mann= 5 ,-1,0
       0      .1       0   325.6    .045       0   381.2      .1       0
     540     .06       0     640      .1       0
Bank Sta=325.6,381.2
XS Rating Curve= 0 ,0
Exp/Cntr(USF)=0,0
Exp/Cntr=0.3,0.1

Type RM Length L Ch R = 1 ,48644   ,243.7,229.7,204.2
XS GIS Cut Line= 4
     2358543.187       705503.712358773.72696762 705334.04190521
 2359024.0071545705164.7480089012359214.37586547704957.475561083
#Sta/Elev= 30
       0 2544.53    11.1 2544.46    70.8 2554.16    94.1 2549.03   105.5 2544.04
   125.4 2529.78   135.3 2517.37   150.2 2505.23   160.2 2489.82   165.1 2484.41
   188.5 2463.47   199.9 2459.88     294 2458.79   390.6 2455.36   432.7 2455.37
     452 2455.58   473.4 2457.96   530.5 2454.72   579.6 2456.33   642.1 2453.25
   663.9 2454.57   674.7  2466.1   696.4    2469   718.4 2484.99   730.6 2487.51
   743.9 2493.62   766.6 2498.53   834.5 2521.22   853.9  2524.3   869.8 2528.98
#Mann= 7 ,-1,0
       0      .1       0   390.6    .045       0   432.7      .1       0
  476.24     .06       0  566.24      .1       0   638.4     .06       0
   768.4      .1       0
Bank Sta=390.6,432.7
XS Rating Curve= 0 ,0
Exp/Cntr=0.3,0.1

Type RM Length L Ch R = 1 ,48414   ,296.9,289.4,275.5
XS GIS Cut Line= 3
2358921.01567838705710.8150800232359064.01215586705328.454933703
2359290.94134839705020.701645201
#Sta/Elev= 30
       0 2534.15    22.4 2525.86    31.6 2524.42    50.3 2517.82   100.1  2505.8
   125.6 2504.49   146.7 2506.77   152.9  2505.6   155.5 2504.52   159.8 2499.78
   181.1 2470.96   202.6 2456.47   223.8 2454.25   255.5 2455.62   270.3 2453.77
   339.4 2453.98   397.3 2457.77   471.9 2455.92   541.5 2457.05     577 2455.87
   601.1 2453.33   619.5 2455.06   630.9 2453.19   640.9 2453.99   650.8  2463.2
   655.8 2466.28     671 2467.61   687.9 2477.69   780.1 2507.16   790.6 2511.71
#Mann= 5 ,-1,0
       0      .1       0   270.3    .045       0   339.4      .1       0
  648.22     .06       0  778.22      .1       0
Bank Sta=270.3,339.4
XS Rating Curve= 0 ,0
Exp/Cntr(USF)=0,0
Exp/Cntr=0.3,0.1

Type RM Length L Ch R = 1 ,48124   ,247.3,252.4,275.4
XS GIS Cut Line= 3
 2359296.9187401705715.2423669272359320.52047463705269.487064078
2359331.54253257705092.724404236
#Sta/Elev= 30
       0  2557.9    18.1 2558.97    26.1 2557.72    49.5 2548.66    90.2 2527.44
   166.3 2497.47   178.3 2490.27   206.7  2469.6   222.4 2460.04   230.4 2456.82
   238.4 2452.16   246.4 2451.29   273.7 2451.22   294.5 2451.66   302.5 2453.08
   326.5 2453.16   338.5 2455.04   422.7 2454.89   458.7 2453.27   474.7 2453.67
   486.8 2452.28   498.8  2453.3   526.8 2451.62   538.9  2452.2   554.9 2463.53
   566.9 2468.31   578.9 2466.14     587 2466.88     611 2479.09   623.5 2483.46
#Mann= 5 ,-1,0
       0      .1       0   246.4    .045       0   294.5      .1       0
  496.38     .06       0  586.38      .1       0
Bank Sta=246.4,294.5
XS Rating Curve= 0 ,0
Exp/Cntr=0.3,0.1

Type RM Length L Ch R = 1 ,47872   ,245.7,249.9,269.6
XS GIS Cut Line= 3
2359479.41544633 705757.185691112359588.52797589 705323.53333004
2359694.84274828704982.206955519
#Sta/Elev= 30
       0 2565.34      33 2552.49    59.9 2536.84      99 2518.05   169.1  2490.9
   189.7 2481.26     205 2471.22   214.8 2457.88   222.7 2451.93   314.6 2449.63
   354.7 2449.54   408.3  2449.8   420.7 2449.99   437.2 2454.85   508.3 2453.07
   529.2 2453.86   580.5 2452.03   600.5 2449.82     613 2452.63   642.4 2454.24
   654.9 2459.28   667.5 2460.21   680.1  2469.5   696.8 2477.89   723.5 2496.93
   734.5 2502.67   755.3 2516.83     768 2522.98   795.7 2543.44   804.7 2547.59
#Mann= 5 ,-1,0
       0      .1       0   314.6    .045       0   408.3      .1       0
  657.17     .06       0  757.17      .1       0
Bank Sta=314.6,408.3
XS Rating Curve= 0 ,0
Exp/Cntr(USF)=0,0
Exp/Cntr=0.3,0.1

Type RM Length L Ch R = 1 ,47622   ,243.2,234.3,225.1
XS GIS Cut Line= 3
2359671.29024322705801.0268019512359711.41135024705689.827768586
2360008.86728839704919.922366927
#Sta/Elev= 30
       0 2573.03    59.4 2541.09   101.9 2515.16   140.4 2485.25   196.1 2455.11
   202.8 2449.66     209 2448.37     269 2448.39   298.7 2450.56   380.5 2451.93
   397.8 2449.56   474.4 2450.25     492 2447.11   513.4 2447.75   530.6 2450.79
   575.4 2447.75   630.9 2447.92   667.8 2453.47   688.4 2454.31   702.1 2451.28
   740.7 2451.06   757.8 2448.18   768.9 2453.77   781.2 2456.33   800.7 2473.89
   822.2  2487.6   830.7 2494.87   865.1 2514.57   907.9 2543.38   943.6 2555.68
#Mann= 5 ,-1,0
       0      .1       0     209    .045       0     269      .1       0
  718.22     .06       0  828.22      .1       0
Bank Sta=209,269
XS Rating Curve= 0 ,0
Exp/Cntr=0.3,0.1

Type RM Length L Ch R = 1 ,47388   ,237.7,257.4,272.4
XS GIS Cut Line= 4
2359873.89920704705779.567748456 2359983.0117366705583.724746682
 2359983.0117366705485.8032457952360248.79866758705024.173313042
#Sta/Elev= 30
       0 2543.86    11.9 2536.19      27 2528.74    38.7 2513.05    43.9 2507.52
    85.2 2484.47   130.9 2456.77   149.3 2451.45   185.5 2452.14   199.6 2447.83
   218.1  2448.3   237.6 2445.72   313.6 2445.42   341.3 2448.06   378.2 2446.68
   475.7 2449.15   496.2 2447.96   510.9 2444.69   539.8 2450.02   566.5 2448.43
   576.7 2445.26   604.6 2449.34   655.2  2449.2   678.2 2447.57   696.7  2448.9
   715.2 2452.92   752.1 2481.94   797.9 2502.15   816.7 2506.72   854.8 2506.78
#Mann= 5 ,-1,0
       0      .1       0   237.6    .045       0   313.6      .1       0
  622.11     .06       0  732.11      .1       0
Bank Sta=237.6,313.6
XS Rating Curve= 0 ,0
Exp/Cntr(USF)=0,0
Exp/Cntr=0.3,0.1

Type RM Length L Ch R = 1 ,47130   ,286.2,303.8,296.5
XS GIS Cut Line= 3
  2359981.145164705922.2199715122360181.44083044705626.888034049
2360558.14038333705087.103208189
#Sta/Elev= 30
       0 2547.25    39.9  2561.9    54.4 2564.14    60.5 2563.77    83.4 2554.16
    90.9 2548.91   106.6 2533.28   131.8 2519.12   190.7 2480.25   198.8 2473.27
   210.3 2459.09   226.3 2443.68   256.4 2445.78   273.6 2442.95   315.4 2445.06
   412.6 2444.11   466.3 2444.08     476 2447.06   549.2  2446.4   568.7 2442.32
   627.2 2447.91   724.9 2447.73   768.7 2445.68   788.2 2448.75   813.9 2470.36
   832.1 2479.81   841.8 2482.77   899.8 2489.78   949.1 2490.37  1015.1 2494.12
#Mann= 5 ,-1,0
       0      .1       0   412.6    .045       0   466.3      .1       0
  726.85     .06       0  886.85      .1       0
Bank Sta=412.6,466.3
XS Rating Curve= 0 ,0
Exp/Cntr=0.3,0.1

Type RM Length L Ch R = 1 ,46827   ,311.5,314.8,322.7
XS GIS Cut Line= 3
2360145.28165236706000.5905647442360360.70895431705740.399148101
2360819.54112989 705323.53333004
#Sta/Elev= 30
       0 2477.88    66.7 2479.83   103.1 2475.92   129.1 2470.35   157.9 2461.69
   169.3 2456.62   186.2 2445.76   206.2  2441.3   227.7 2440.13   255.4 2441.44
   299.3 2445.02   336.8 2442.53   365.2 2442.78   380.3  2444.6   455.6 2443.18
   499.2 2444.47   523.8 2444.11   544.8 2440.44   556.7 2443.18   574.9 2443.57
   591.1 2440.24   623.5  2446.1   747.5 2445.44     753 2446.41   769.4 2455.71
   785.6 2461.74   861.3 2472.05   937.4 2485.53   947.8  2489.3   957.7 2490.81
#Mann= 5 ,-1,0
       0      .1       0   206.2    .045       0   255.4      .1       0
   637.8     .06       0   767.8      .1       0
Bank Sta=206.2,255.4
XS Rating Curve= 0 ,0
Exp/Cntr(USF)=0,0
Exp/Cntr=0.3,0.1

Type RM Length L Ch R = 1 ,46512   ,116.9,120,125.5
XS GIS Cut Line= 3
2360290.62727325706208.8678158142360400.57006348706126.299126019
2360987.53375815705697.475950986
#Sta/Elev= 30
       0 2464.92    26.9 2462.23      47 2457.95     153 2457.15   196.5  2455.7
   216.3 2452.66   220.8 2449.91   227.5 2442.29   232.5 2439.45   258.2 2440.33
   275.4 2439.29   321.2 2439.21   345.1 2441.74   369.8 2440.59   381.3 2441.49
   397.1 2440.09     410 2440.69   415.7 2439.37   435.7 2438.25   464.9 2440.34
   501.6 2439.13   513.5 2439.77   528.4 2442.77   630.4 2445.38   711.6 2449.22
   746.3 2448.84     786 2450.61   802.1 2455.42   817.5  2464.5   864.4 2477.71
#Mann= 5 ,-1,0
       0      .1       0   275.4    .045       0   321.2      .1       0
   727.5     .06       0   827.5      .1       0
Bank Sta=275.4,321.2
XS Rating Curve= 0 ,0
Exp/Cntr=0.3,0.1

Type RM Length L Ch R = 1 ,46392   ,261.8,276,284.6
XS GIS Cut Line= 3
2360308.72897175706274.1466276032360817.92077636706025.146239634
 2361184.4269654705974.786610606
#Sta/Elev= 30
       0 2470.13    21.6 2466.29   150.8 2455.97   181.9 2454.79   226.5  2455.9
   230.6 2454.32   245.5 2440.87   251.5 2437.94   275.4 2439.94   284.4 2438.47
   342.2 2438.68   364.5 2440.87     404 2441.38   440.2 2437.12   457.8 2439.11
   480.3 2439.61   515.9 2436.92   541.6 2438.42   560.4  2441.3   585.2 2439.55
   617.5 2441.24   698.3 2439.23   738.7 2441.79   746.7 2440.65   771.1 2441.34
   803.3 2440.04   815.4 2446.23   827.9  2456.8   908.2 2518.12   936.8 2536.91
#Mann= 5 ,-1,0
       0      .1       0   284.4    .045       0   342.2      .1       0
  726.81     .06       0  826.81      .1       0
Bank Sta=284.4,342.2
XS Rating Curve= 0 ,0
Exp/Cntr(USF)=0,0
Exp/Cntr=0.3,0.1

Type RM Length L Ch R = 1 ,46116   ,238.2,224.9,220.2
XS GIS Cut Line= 3
 2360317.6678082706415.3692147322360580.50670049 706383.88103961
2361305.50283786706320.730158192
#Sta/Elev= 30
       0 2477.43     208 2453.51   224.1 2449.33   240.2  2437.4   248.3  2435.7
   318.6 2435.81   318.6 2435.82   328.6 2437.62   380.8 2435.44   412.9 2437.45
   441.1  2434.3   469.2  2438.2   501.3 2434.96   533.4 2436.94   549.5 2433.39
   573.6 2435.41   649.8  2435.3     699 2438.35   730.1 2435.75   746.2 2440.96
   758.2 2441.68   762.3    2443   774.3 2455.01   790.4 2465.76   802.5  2470.9
   822.5 2484.39   830.5 2487.04   882.7 2522.25   922.9 2546.94   992.5 2570.86
#Mann= 5 ,-1,0
       0      .1       0   248.3    .045       0   318.6      .1       0
  764.72     .06       0  864.72      .1       0
Bank Sta=248.3,318.6
XS Rating Curve= 0 ,0
Exp/Cntr=0.3,0.1

Type RM Length L Ch R = 1 ,45891   ,252.6,250.9,257
XS GIS Cut Line= 4
2360324.92666082706608.6160584922360627.04058232706614.541988842
2360756.79152974706567.3432066872361199.40508589706584.760464345
#Sta/Elev= 30
       0 2504.68    59.3 2484.29    75.3  2480.7    87.3 2475.73    99.3  2474.4
   111.3 2470.49   159.3 2461.25   255.3 2447.53   291.3 2436.51   303.4 2435.17
   322.8 2435.85   338.5 2433.66   401.3 2433.27     414  2435.6   447.6 2433.93
   471.6 2435.66   515.7 2435.22   547.7 2431.42   571.7 2435.24   635.8 2432.03
   659.8 2434.31   723.8 2431.99   755.9 2437.04   767.9 2442.87   783.9 2443.92
   788.1 2447.74   799.9 2464.84   823.9 2484.27   855.9 2504.93   883.2 2517.59
#Mann= 5 ,-1,0
       0      .1       0   338.5    .045       0   401.3      .1       0
  660.24     .06       0  860.24      .1       0
Bank Sta=338.5,401.3
XS Rating Curve= 0 ,0
Exp/Cntr(USF)=0,0
Exp/Cntr=0.3,0.1

Type RM Length L Ch R = 1 ,45640   ,155.8,155.1,152.9
XS GIS Cut Line= 4
     2360347.754      706930.7122360643.96607457706857.922775822
2360912.38276303706791.0590473942361197.23480924706766.424000591
#Sta/Elev= 30
       0 2512.37    44.6 2488.81    58.1 2479.85    67.7 2471.59    78.7 2468.62
   111.6 2445.22     124 2438.55   132.2 2435.89   165.2 2433.44     194 2434.87
   210.5 2431.74   222.9 2431.13   239.3 2433.52   309.8 2434.66   338.2 2431.03
   408.3 2432.94   444.4 2430.99     499 2430.42   519.6 2433.94   540.2 2435.46
   589.5 2432.08   605.7 2433.37   621.6 2429.61   697.9 2432.94   717.9 2447.64
     734 2449.16   758.1 2469.35   777.1 2479.17   830.4 2497.92   867.6 2505.19
#Mann= 5 ,-1,0
       0      .1       0   444.4    .045       0     499      .1       0
  651.64     .06       0  741.64      .1       0
#XS Ineff= 2 , 0
          189.37  2444.5
Permanent Ineff=
       F       F
Bank Sta=444.4,499
XS Rating Curve= 0 ,0
Exp/Cntr=0.3,0.1

Type RM Length L Ch R = 1 ,45485   ,247.3,244.1,239.9
XS GIS Cut Line= 2
2360436.87962025707094.1514949562361103.28440769706885.479288787
#Sta/Elev= 30
       0 2487.36      13 2477.53    32.1 2460.07    45.4 2455.45    62.1 2442.07
      80  2431.5    92.8 2430.08   112.4 2432.31   246.6 2432.85   259.1 2432.45
   275.9  2428.3   368.1 2431.42   397.5 2429.19   447.1 2429.47   464.5 2433.03
   485.4 2433.81   498.1 2433.21   510.6 2429.92   523.2 2431.86   544.2 2429.52
   560.9 2431.19   577.7 2428.77   602.8  2429.9   615.4 2434.44   632.2 2447.83
   648.9 2450.99   653.1 2453.54   661.5 2462.95   665.7 2465.83   698.3  2472.2
#Mann= 5 ,-1,0
       0      .1       0   397.5    .045       0   447.1      .1       0
     570     .06       0     670      .1       0
Bank Sta=397.5,447.1
XS Rating Curve= 0 ,0
Exp/Cntr(USF)=0,0
Exp/Cntr=0.3,0.1

Type RM Length L Ch R = 1 ,45241   ,149.3,150.7,142.4
XS GIS Cut Line= 2
2360487.13113639707408.1797978792361029.23578316707143.107942157
#Sta/Elev= 30
       0 2532.81    14.5 2524.46    71.8  2494.5   130.3 2468.71   152.5  2456.1
   161.5 2449.34   183.7 2436.12   197.1 2432.42   224.3 2429.12   237.1 2431.11
   286.1 2432.31   293.1 2431.75   303.9 2428.54     311 2427.69     317 2427.65
   339.6  2430.4   361.7 2429.79   370.8 2427.66   410.8 2429.69   433.1 2426.54
   455.3  2428.7   464.2 2426.56   486.5 2426.26   508.8 2426.98   514.4 2428.91
   517.7  2431.7   522.1 2436.87   526.3 2439.93     531 2441.15   603.4 2443.38
#Mann= 3 ,-1,0
       0      .1       0   464.2    .045       0   508.8      .1       0
Bank Sta=464.2,508.8
XS Rating Curve= 0 ,0
Exp/Cntr(USF)=0,0
Exp/Cntr=0.3,0.1

Type RM Length L Ch R = 1 ,45090   ,235,222.4,202.2
XS GIS Cut Line= 3
2360559.70076244707572.6397162282361016.31909597707302.167476303
 2361195.9800942707024.530143955
#Sta/Elev= 30
       0 2573.72    14.5 2565.73    79.6 2524.88   124.5 2498.48     140 2487.97
   204.3 2453.29     251 2429.49   256.2 2427.65   262.7    2427   277.3 2430.14
     305 2429.95   316.7  2426.4     326 2425.81   338.6 2428.74   353.2 2429.64
   370.7 2426.95   391.1 2428.24   436.2 2425.87   493.4 2426.41   516.6 2426.86
   536.7  2426.1   548.7  2428.9   574.6 2430.66     595 2435.18   713.6 2444.65
   741.5 2448.79   759.8 2452.88   771.4 2448.78   788.1    2452   861.4 2455.03
#Mann= 4 ,-1,0
       0      .1       0   436.2    .045       0   493.4      .1       0
  780.71     .06       0
Bank Sta=436.2,493.4
XS Rating Curve= 0 ,0
Exp/Cntr=0.3,0.1

Type RM Length L Ch R = 1 ,44868   ,294.4,296.1,279.6
XS GIS Cut Line= 3
2360927.52073711707888.106775204 2361095.3861672707370.521699088
2361285.63365464707018.004295895
#Sta/Elev= 30
       0 2721.96    40.9 2705.52    53.5 2697.72    57.7 2692.87    79.9 2655.23
   116.6 2628.48   155.3 2606.83   162.9 2598.05   171.3 2582.66   183.9 2573.44
   196.6 2557.06   225.9 2527.26   255.4 2500.71   269.6  2484.8     289 2461.76
   297.4 2441.85   318.5 2428.48   335.3 2424.93   356.3 2425.16   402.9 2424.45
   474.1 2425.88   516.1 2423.29   537.1 2427.16   604.7 2430.06   677.5 2429.12
   700.2 2434.96   786.6 2450.25   802.5 2446.71   814.3 2449.42   944.7 2454.61
#Mann= 5 ,-1,0
       0      .1       0   356.3    .045       0   402.9      .1       0
  744.13     .06       0  914.13      .1       0
Bank Sta=356.3,402.9
XS Rating Curve= 0 ,0
Exp/Cntr(USF)=0,0
Exp/Cntr=0.3,0.1

Type RM Length L Ch R = 1 ,44572   ,244.3,247.2,241.7
XS GIS Cut Line= 2
     2361323.276      707922.0572361262.95353985707117.173561535
#Sta/Elev= 30
       0 2560.24    85.1 2553.26   181.4 2540.22   245.6 2526.97   297.7 2511.46
   337.8  2493.4   349.9 2485.42   361.9 2471.25   365.9 2465.08   369.9 2454.14
   373.9 2438.46   377.9 2429.84     394 2423.08   413.9 2421.63   454.1 2424.93
   498.3 2422.87   511.2 2421.76   554.4 2423.12   566.5    2427   622.6 2425.88
   654.7 2428.69     687 2426.85   694.8 2428.43   706.9 2433.96   714.9 2435.21
   730.9  2442.1     751  2448.3     763 2444.72     775  2447.9   807.1 2449.64
#Mann= 4 ,-1,0
       0      .1       0   498.3    .045       0   554.4      .1       0
     730     .06       0
Bank Sta=498.3,554.4
XS Rating Curve= 0 ,0
Exp/Cntr=0.3,0.1

Type RM Length L Ch R = 1 ,44324   ,181.6,177.1,174.6
XS GIS Cut Line= 3
2361576.60040013707804.174060158 2361509.4542281707345.341884574
2361492.66768509707018.004295895
#Sta/Elev= 30
       0 2473.81   176.9 2475.77   214.6 2473.52   298.1 2462.63   310.3 2460.07
   322.4 2455.42   326.4  2451.7   330.5 2444.04   334.5 2434.66   342.6 2423.77
   346.6 2421.01   353.5 2420.49   399.2 2419.79   405.6 2420.35   423.5 2424.13
   455.8  2423.2   479.9 2424.04   499.9 2422.33   511.9  2424.9     540  2422.3
     576 2424.25   608.1 2421.95   632.1 2425.92   652.1 2434.53   668.2 2438.64
   680.2 2438.89   692.2 2441.87   728.2 2445.54   760.3 2447.16   791.5 2450.65
#Mann= 5 ,-1,0
       0      .1       0   353.5    .045       0   405.6      .1       0
  513.72     .06       0  613.72      .1       0
Bank Sta=353.5,405.6
XS Rating Curve= 0 ,0
Exp/Cntr(USF)=0,0
Exp/Cntr=0.3,0.1

Type RM Length L Ch R = 1 ,44147   ,280.8,304,312
XS GIS Cut Line= 3
2361695.19028791707607.111235196 2361700.2944763707416.963905212
2361581.33466706706990.308571682
#Sta/Elev= 30
       0 2449.34      82 2448.85     110 2446.16     130 2442.48     146 2437.04
   162.6 2426.03     174 2421.62   205.6 2422.17   231.5 2419.12   238.8    2419
   281.3 2419.11   302.1 2421.48   351.9 2422.92   368.6 2420.43   381.7 2422.85
   405.9 2423.62   430.4 2422.95   439.1 2421.25   459.9 2421.82   468.2 2425.41
   484.8 2436.17   501.9 2436.54   505.6 2437.05   513.9 2441.82   538.8 2444.87
   555.4 2445.17     572 2448.87   584.5 2449.78   617.7 2456.72   633.1 2461.94
#Mann= 5 ,-1,0
       0      .1       0   231.5    .045       0   281.3      .1       0
  420.22     .06       0  520.22      .1       0
Bank Sta=231.5,281.3
XS Rating Curve= 0 ,0
Exp/Cntr=0.3,0.1

Type RM Length L Ch R = 1 ,43843   ,188.1,192,192.9
XS GIS Cut Line= 3
 2361764.0501304707619.5220870572361926.32004616707378.914970592
2362096.98323342706984.431209876
#Sta/Elev= 30
       0 2443.72    94.5  2441.6   164.8  2436.1     191 2432.36   195.8  2430.7
   210.3    2422   229.6 2416.94   248.9 2419.14   277.8 2419.57   292.1 2421.13
   317.3  2419.4   344.4  2420.4   355.3 2416.88   362.9 2416.13   384.2 2415.49
   408.5 2416.02   418.5 2418.45   431.6  2426.8     449 2428.92   475.2 2453.96
   492.6  2462.4   502.9 2469.87   563.7 2503.69   592.8 2524.63   610.3 2529.94
   627.6 2530.99   645.1 2535.05   684.3 2535.23   710.5 2532.28     720 2533.95
#Mann= 4 ,-1,0
       0      .1       0   362.9    .045       0   408.5     .06       0
  490.21      .1       0
Bank Sta=362.9,408.5
XS Rating Curve= 0 ,0
Exp/Cntr(USF)=0,0
Exp/Cntr=0.3,0.1

Type RM Length L Ch R = 1 ,43651   ,266.1,266.6,280.4
XS GIS Cut Line= 5
2361854.10561808707649.1746472792362014.33239249707575.994251505
2362093.05147571707451.9717150462362211.31299319707234.050207087
      2362317.92      707019.444
#Sta/Elev= 30
       0 2440.02    59.4 2435.73   143.4 2436.32   156.2 2435.15   169.4 2436.76
   217.2 2434.69   231.2 2432.82   239.3 2429.99   255.3 2420.05   263.6 2416.96
   293.2 2417.12   307.4 2413.77   368.7 2417.92   381.9 2417.17   395.3  2415.4
   413.5 2416.64   433.6 2417.97   444.5 2416.97   453.6 2422.35   471.9 2428.78
   489.7 2444.75   508.3 2457.75   564.4 2492.17   589.8 2511.21   603.2 2518.35
   612.2 2525.58   656.8 2546.01   679.2 2552.49   727.4 2560.05   810.6 2579.66
#Mann= 4 ,-1,0
       0      .1       0   381.9    .045       0   413.5     .06       0
  503.04      .1       0
Bank Sta=381.9,413.5
XS Rating Curve= 0 ,0
Exp/Cntr=0.3,0.1

Type RM Length L Ch R = 1 ,43385   ,240.4,241,251.9
XS GIS Cut Line= 4
2361984.95954207707712.203590106   2362163.76367707666.006606334
2362292.82623519707560.7691865252362586.59073785707297.780012714
#Sta/Elev= 30
       0 2431.94      57 2432.03    90.1  2434.1   126.6 2432.91   188.4 2433.85
   195.5 2431.89   205.5 2421.23   216.8 2413.59   236.7  2414.1   257.5 2412.32
   268.3 2412.46   296.4 2415.69   333.4 2415.46   377.2 2417.03   392.6 2415.08
   415.6  2416.4   450.6 2414.27   489.9 2414.12   514.8 2416.62   524.5 2420.68
   540.2 2423.55   551.6 2429.58   562.9 2433.96   602.5 2455.64   632.4 2473.44
   662.4 2486.41   679.1 2488.16   715.4 2482.41   731.5 2481.46   745.5 2482.08
#Mann= 4 ,-1,0
       0      .1       0   450.6    .045       0   489.9     .06       0
  601.21      .1       0
Bank Sta=450.6,489.9
XS Rating Curve= 0 ,0
Exp/Cntr(USF)=0,0
Exp/Cntr=0.3,0.1

Type RM Length L Ch R = 1 ,43144   ,229.5,227.5,243.6
XS GIS Cut Line= 3
2361744.61628673707888.1537606662362590.56452043707641.279306012
2362733.93066529707560.795238152
#Sta/Elev= 30
       0 2453.72    45.4 2446.89    98.8 2442.03   157.9 2438.96   257.9 2430.85
   345.4 2429.05   382.7 2431.92   470.4 2432.06   482.9 2429.11   495.4 2414.14
   503.7 2411.27   520.4  2411.2   545.4 2414.14   628.7 2414.66   647.2 2414.04
   657.9  2411.5   670.4 2414.28   682.9 2414.53   703.7 2410.76   720.4 2413.38
   782.6 2414.36   803.7 2414.13   824.5 2411.16   853.6 2411.56   870.4 2412.36
   894.2 2416.88     929  2417.3   942.7 2421.16   979.4  2426.5  1045.6 2427.95
#Mann= 4 ,-1,0
       0      .1       0   824.5    .045       0   853.6     .06       0
  951.24      .1       0
Bank Sta=824.5,853.6
XS Rating Curve= 0 ,0
Exp/Cntr=0.3,0.1

Type RM Length L Ch R = 1 ,42916   ,290.8,301,306.3
XS GIS Cut Line= 5
2361702.71078972707947.8757106112362106.83126957707889.157350291
2362414.23915595707854.6171383382362562.76206735  707882.2493079
2362908.16418688707923.697562244
#Sta/Elev= 30
       0 2463.06    70.2 2451.92    81.3 2451.89   191.5 2439.33   203.6 2439.48
   284.4 2431.67   393.6 2426.36   441.9 2428.93   490.2 2427.54   494.2  2426.1
   503.6 2416.13   514.2 2412.12   534.5 2412.44   570.7 2410.08   594.9 2412.07
     611 2409.51   636.6 2412.57   679.4 2409.64   731.7 2412.78   746.9 2410.45
   772.6 2410.32   810.8 2415.33   914.5  2412.5   991.1 2416.89  1003.1 2415.29
  1099.3 2415.66    1120 2424.28    1164 2424.73  1196.5 2428.99  1216.7 2429.54
#Mann= 5 ,-1,0
       0      .1       0   746.9    .045       0   772.6      .1       0
  857.71     .06       0  958.78      .1       0
#XS Ineff= 2 , 0
                          990.84         2421.98
Permanent Ineff=
       F       F
Bank Sta=746.9,772.6
XS Rating Curve= 0 ,0
Exp/Cntr(USF)=0,0
Exp/Cntr=0.3,0.1

Type RM Length L Ch R = 1 ,42615   ,149.9,148.9,142.9
XS GIS Cut Line= 3
 2361834.2636646708004.1629673332362131.59867643707915.504064635
2362362.76926349708203.030676023
#Sta/Elev= 30
       0 2445.52    35.4 2439.93    52.1 2435.17    60.4 2434.04      73 2433.63
    89.6 2435.01   135.8 2433.09   198.2 2427.82   277.2 2426.98   298.4 2424.93
   317.5 2425.88   343.2 2422.19   348.9 2420.31   358.6 2414.58   368.9 2410.92
   399.7 2408.44   417.1 2408.43   451.6 2408.53   486.9 2408.33   521.9 2409.71
   533.1  2408.3   562.2  2411.4   592.1 2408.16     624 2407.97   639.1 2406.64
   649.5 2407.12   656.1 2409.12   661.8 2415.67     676 2437.62   679.2 2441.51
#Mann= 3 ,-1,0
       0      .1       0   417.1    .045       0   451.6      .1       0
Bank Sta=417.1,451.6
XS Rating Curve= 0 ,0
Exp/Cntr=0.3,0.1

Type RM Length L Ch R = 1 ,42466   ,371.3,336.3,309.2
XS GIS Cut Line= 5
2361711.76638265708078.5741116452361977.45647764708012.314877157
2362252.67671425708220.1843950842362310.93162216708221.075735104
2362593.56844267708152.352481514
#Sta/Elev= 30
       0 2464.09    66.4 2451.24     120 2445.38   169.4 2437.75   281.9 2425.79
   312.3 2417.05   327.8 2410.39   365.3 2411.54   373.5 2409.97   407.6 2407.95
   436.3 2407.73   454.5 2406.69   482.8 2410.01   516.3 2410.03   550.5 2407.46
   557.9 2405.86   626.2 2424.36   645.6 2427.54   690.6 2432.31   715.3 2437.67
   765.8 2455.17   793.5 2461.76   830.6 2468.74   851.2  2468.4   879.9 2460.14
   908.8 2456.37     923 2451.18   937.6 2449.93   962.3 2441.87   967.9 2441.34
#Mann= 3 ,-1,0
       0      .1       0   407.6    .045       0   436.3      .1       0
Bank Sta=407.6,436.3
XS Rating Curve= 0 ,0
Exp/Cntr(USF)=0,0
Exp/Cntr=0.3,0.1

Type RM Length L Ch R = 1 ,42130   ,200.3,194.2,192.3
XS GIS Cut Line= 3
2361613.21331539 708697.879526622362169.12563194708309.021631366
2362622.07465712708183.764447627
#Sta/Elev= 30
       0 2535.75    13.4 2526.37    42.7 2509.58    81.7 2482.56    91.5 2478.95
   147.8  2437.3   171.6 2417.47   189.1  2408.6   247.7 2405.73   315.3 2408.04
   403.9 2408.05   423.4 2404.97   467.4 2406.52   485.2 2404.82   490.9 2404.47
   548.4 2405.13   628.4 2407.52   664.2 2404.81     723 2409.91     748 2409.52
   768.5 2419.19   791.3 2425.82   859.6 2433.07   934.7 2453.65   984.5  2463.9
  1013.6 2463.07  1064.4 2453.25  1084.1 2451.41  1138.1 2436.49  1148.4  2436.2
#Mann= 3 ,-1,0
       0      .1       0   485.2    .045       0   548.4      .1       0
Bank Sta=485.2,548.4
XS Rating Curve= 0 ,0
Exp/Cntr=0.3,0.1

Type RM Length L Ch R = 1 ,41936   ,570.5,558.7,533.2
XS GIS Cut Line= 3
2361744.72280638708867.3258775122362479.11688769708289.286665129
2362635.47175661708213.478243833
#Sta/Elev= 30
       0 2529.62    90.9 2472.61   132.2 2440.41   157.1  2417.7   171.6    2408
   182.6 2405.17     208 2407.73   234.7 2405.98   243.6 2403.53   268.6 2402.96
   294.5 2406.69   311.6 2405.17   365.7 2406.88   414.2  2404.7   467.6 2406.46
   536.6 2404.42   579.1 2404.05   625.4 2407.63   696.2 2406.88     736 2404.35
   760.1 2416.27   781.6 2423.95   844.3 2433.79   863.6 2439.09   876.6 2445.01
   889.8 2445.28   935.5 2454.54  1022.3 2450.38  1049.2 2446.57  1108.4 2432.94
#Mann= 3 ,-1,0
       0      .1       0   536.6    .045       0   579.1      .1       0
Bank Sta=536.6,579.1
XS Rating Curve= 0 ,0
Exp/Cntr(USF)=0,0
Exp/Cntr=0.3,0.1
