HEC-RAS study GLADYFK.prj: GLADYFK

--- GLADYFK.g01 (geometry) --- (continued)

Type RM Length L Ch R = 1 ,41377   ,310.7,307,301.4
XS GIS Cut Line= 4
2362382.21338303 709230.714286972362384.47956634708838.664574991
2362454.22948409708439.7608603472362490.17453167708389.783197634
#Sta/Elev= 30
       0  2527.3    57.5 2493.87    85.5 2483.02    97.5 2475.56   113.5  2473.8
   125.5 2466.78   146.7 2459.11   186.4 2437.47   225.5 2422.33   233.5 2416.15
   241.5 2403.68   249.5 2399.81   257.5 2399.93   297.8 2400.86   341.5 2401.94
   369.7 2399.25   389.5 2399.56   417.3 2403.04   451.8 2401.25   470.7 2402.94
     491 2399.26   503.2 2403.02   515.4 2403.55   592.5 2402.08   726.5 2404.19
   742.8 2402.05     759  2407.6   779.3  2419.1   800.2  2427.3   858.6 2442.75
#Mann= 3 ,-1,0
       0      .1       0   257.5    .045       0   297.8      .1       0
Bank Sta=257.5,297.8
XS Rating Curve= 0 ,0
Exp/Cntr(USF)=0,0
Exp/Cntr=0.3,0.1

Type RM Length L Ch R = 1 ,41070   ,211.7,210,206.4
XS GIS Cut Line= 4
2362729.45183306709153.8599645292362652.58570322708769.236853237
2362655.31762451708478.7253557992362634.33984107 708378.47727202
#Sta/Elev= 30
       0 2483.81    61.9 2459.41    94.5 2448.49   110.8 2446.97   131.2 2441.45
   196.5 2431.21   229.1 2423.79   237.3 2420.18   253.6 2406.41   264.3 2400.38
     274 2398.14   300.8 2397.95   335.7 2397.57   355.2  2399.7   380.1 2399.91
   388.2  2397.7   404.3 2396.34   440.3  2402.1   480.3 2400.88   550.4 2402.86
   572.3  2400.9   596.3 2403.57   620.3 2401.85   632.3 2402.75   637.6 2404.25
   651.1 2414.94   664.3 2421.67   704.8 2434.42   737.4 2438.64   785.2 2439.06
#Mann= 3 ,-1,0
       0      .1       0   300.8    .045       0   335.7      .1       0
Bank Sta=300.8,335.7
XS Rating Curve= 0 ,0
Exp/Cntr=0.3,0.1

Type RM Length L Ch R = 1 ,40860   ,203.6,216.6,220.2
XS GIS Cut Line= 5
2362769.99948211 709064.855292472362858.11117345708916.004685715
2362872.35950854708800.7228017192362826.27228713708671.684730122
2362856.96341477708390.635294286
#Sta/Elev= 30
       0 2450.71     8.9 2447.22    39.3 2444.35    60.1 2443.63   132.7  2445.7
   162.3 2443.43     167 2440.04   183.9 2408.18   187.9 2402.95   212.1 2395.78
   228.2 2395.66   240.3 2399.88   298.3  2399.2   331.1 2396.48     364 2396.68
   399.1 2395.04     411 2395.73   426.8 2400.75   472.9 2400.76     489 2399.48
   545.4 2401.89   565.5 2409.07   581.6 2418.57   597.7 2422.93   636.9  2424.4
     654 2422.26   662.1 2423.94   673.2  2428.5   694.2 2426.89   708.9 2428.05
#Mann= 4 ,-1,0
       0      .1       0   331.1    .045       0     364      .1       0
  526.15     .06       0
Bank Sta=331.1,364
XS Rating Curve= 0 ,0
Exp/Cntr(USF)=0,0
Exp/Cntr=0.3,0.1

Type RM Length L Ch R = 1 ,40643   ,696.1,748.3,782
XS GIS Cut Line= 4
2362833.82099452709073.6706962942362931.24919236709010.085073416
2363100.87950189708517.8542645122363093.79409033  708226.4797212
#Sta/Elev= 30
       0 2432.84    45.8 2420.86   112.7 2410.21   152.4 2399.86   218.8 2399.22
   265.4 2394.47   278.1 2398.28   307.7 2399.01   328.8 2394.16   391.5 2397.82
   462.9 2394.91   489.6 2395.06     515 2397.93   548.9 2396.78   578.5 2399.39
   591.2  2403.4   603.8 2412.92     625 2414.36     650 2426.72   665.7 2432.34
   681.7 2434.95   697.7 2441.88   709.7 2442.14   757.7 2451.29   769.7 2455.45
   796.9 2458.56   845.7 2470.05   865.7 2472.72   909.7 2466.33   928.4  2466.7
#Mann= 5 ,-1,0
       0      .1       0   462.9    .045       0   489.6      .1       0
  576.34     .06       0  686.98      .1       0
Bank Sta=462.9,489.6
XS Rating Curve= 0 ,0
Exp/Cntr=0.3,0.1

Type RM Length L Ch R = 1 ,39895   ,326.9,323.5,314.8
XS GIS Cut Line= 4
2362807.57266272709130.3601277292362982.74410775709134.278692893
2363498.90925911708982.0792770822363971.41554047709036.883172946
#Sta/Elev= 30
       0  2444.7    16.6 2440.62    24.6 2436.24    60.6 2422.72    92.6 2414.68
   116.6  2410.3   177.3 2404.15   214.2 2395.92   301.8 2396.79   318.5 2395.32
   351.9 2396.73   401.9 2391.87   451.9 2395.21   489.5 2393.54   702.2 2395.13
   713.4 2394.28   722.7 2390.77   742.5 2388.47   787.22390.116   795.2 2398.25
   811.3 2401.16   829.1 2425.95   839.5  2437.5   847.5 2444.28   867.6 2457.21
   936.1 2495.05   976.4 2519.32  1056.9 2554.79  1113.3 2576.55    1189 2598.76
#Mann= 4 ,-1,0
       0      .1       0   722.7    .045       0   787.2     .06       0
  853.35      .1       0
Bank Sta=722.7,787.2
XS Rating Curve= 0 ,0
Exp/Cntr=0.3,0.1

Type RM Length L Ch R = 1 ,39572   ,255.8,242.3,227.4
XS GIS Cut Line= 5
2362906.34556672709471.5106978112363109.35535019709326.805019843
2363306.29495219 709288.854134692363709.17198441709291.651891858
2363829.43715681709278.349527786
#Sta/Elev= 30
       0 2423.86    11.6 2423.97    61.2 2415.38   125.1  2407.3   134.9 2407.16
   213.5 2395.68   256.5 2394.28   292.9 2391.35   301.1 2393.31   333.6  2393.2
   345.9 2391.02   370.3 2392.15   382.5 2390.72   427.3 2392.55   447.7 2387.16
   467.7 2386.72   523.7 2392.12     528 2392.16   539.42388.548   560.2 2387.01
   619.8 2387.44   643.8 2390.99   651.8 2393.53   663.8 2394.38   667.8 2396.02
     681  2406.8   739.8 2437.55   795.8 2461.07   912.1 2507.26   973.8  2526.5
#Mann= 5 ,-1,0
       0      .1       0   539.4    .045       0   619.8      .1       0
  679.87     .06       0  779.87      .1       0
Bank Sta=539.4,619.8
XS Rating Curve= 0 ,0
Exp/Cntr=0.3,0.1

Type RM Length L Ch R = 1 ,39329   ,183.6,182,180.8
XS GIS Cut Line= 2
2362864.66125114 709669.624257292363850.09349816709420.934731228
#Sta/Elev= 30
       0 2464.13      82  2428.5   144.9 2405.94   184.4  2404.4   197.6 2401.18
   250.3 2394.51   273.4 2389.62     313 2386.16   355.7 2386.84   383.2 2388.79
   421.6 2389.17   440.9 2387.59   454.6 2389.54   490.4 2390.11   502.8 2389.33
   519.3 2385.69   597.7 2386.08   618.3 2384.74   626.6 2385.75   655.7  2389.3
   729.7 2390.77   733.8 2392.39   746.2 2402.69   762.7 2410.67   783.3 2423.13
   791.6 2425.01   808.1 2435.25   845.2 2449.92   894.7 2464.92  1016.3 2495.33
#Mann= 5 ,-1,0
       0      .1       0   519.3    .045       0   626.6      .1       0
     690     .06       0     800      .1       0
Bank Sta=519.3,626.6
XS Rating Curve= 0 ,0
Exp/Cntr(USF)=0,0
Exp/Cntr=0.3,0.1

Type RM Length L Ch R = 1 ,39147   ,234.5,225.8,215.5
XS GIS Cut Line= 3
2362845.07554289709870.1044172652363787.38171555709619.195165469
2363929.19001328709577.855596016
#Sta/Elev= 30
       0  2540.3    49.1    2508    65.4 2494.86    81.9 2486.66   123.2 2459.79
   135.7 2455.27   156.4 2439.88   168.8 2436.46     235  2392.8   247.4 2391.77
     264 2386.59   288.8 2384.49   342.6 2387.14   425.4 2385.14     442 2387.52
   516.5 2389.28   566.2 2387.75     608 2383.57   690.3 2383.12   694.5 2384.46
   702.8 2387.47   715.2 2387.84   814.5 2384.32   831.1 2386.66   847.6 2397.39
   872.8 2409.55   922.1 2428.97  1054.8 2437.97  1096.8 2442.88  1122.9 2448.78
#Mann= 5 ,-1,0
       0      .1       0     608    .045       0   694.5      .1       0
     820     .06       0     830      .1       0
Bank Sta=608,694.5
XS Rating Curve= 0 ,0
Exp/Cntr=0.3,0.1

Type RM Length L Ch R = 1 ,38921   ,280.6,280.9,278.4
XS GIS Cut Line= 3
2363038.74391938710185.6550238682363700.87978252709828.163830154
2363915.37449875709710.036305275
#Sta/Elev= 30
       0 2452.61    24.4 2445.73    36.8 2439.46    56.2 2432.14    93.6 2422.92
    98.8  2419.8   110.7 2406.94   131.3 2390.26     138 2386.34   154.9 2382.48
   199.2 2383.72   215.3 2385.57   287.7 2383.24   314.3  2385.9   361.5 2386.38
   456.2 2384.69   483.5 2385.65   510.8  2384.9     521 2382.36   556.2 2381.47
   601.7 2381.65   624.4 2384.75   647.1 2385.91   768.9 2383.35   800.1  2384.6
   833.7 2383.59   865.8 2399.99   910.2 2411.96   934.3 2415.44   997.4 2417.67
#Mann= 5 ,-1,0
       0      .1       0     521    .045       0   601.7      .1       0
  792.48     .06       0  902.48      .1       0
Bank Sta=521,601.7
XS Rating Curve= 0 ,0
Exp/Cntr(USF)=0,0
Exp/Cntr=0.3,0.1

Type RM Length L Ch R = 1 ,38641   ,239.2,235,223.9
XS GIS Cut Line= 3
2363152.71978141710461.1684637492363793.57191379710088.797635427
2363986.50102276 709777.22872116
#Sta/Elev= 30
       0 2484.78    63.7 2480.75     152 2472.27   191.1 2462.72   207.6 2456.89
   263.1 2430.31   294.6 2405.09   310.5 2389.27   318.5 2384.56   327.8 2382.48
   350.3 2380.89   420.4 2380.87   494.4 2384.13   512.9 2380.99   540.6 2380.11
   546.8 2380.02   614.7 2380.32   660.9 2380.57   698.9 2383.23   730.3 2381.27
   784.1 2384.48   820.7 2381.66   839.5 2383.97   870.6 2384.39   886.6 2381.76
   914.8  2383.5   949.1    2381   991.4 2381.59  1036.3 2393.14  1107.6 2403.95
#Mann= 5 ,-1,0
       0      .1       0   540.6    .045       0   614.7      .1       0
  901.18     .06       0 1021.18      .1       0
Bank Sta=540.6,614.7
XS Rating Curve= 0 ,0
Exp/Cntr=0.3,0.1

Type RM Length L Ch R = 1 ,38406   ,272.6,267.7,268.5
XS GIS Cut Line= 3
2363480.16782814710760.7495528872363756.83492589710303.782548748
2364151.62954851709834.381068306
#Sta/Elev= 30
       0 2450.56   139.8 2468.57   228.6 2476.99   293.5 2478.25   303.4 2475.76
   345.5 2452.94   368.9 2409.18   378.3 2402.23   393.9 2394.78     411 2378.99
   415.7 2377.81   432.5 2377.32   462.4 2377.96   471.8 2381.15   503.6 2378.23
   542.8 2381.93   579.4 2378.78   717.3 2377.88     731 2382.13   741.4 2382.51
     778 2380.04   812.8 2381.82   836.5 2379.57   881.2 2384.84   945.3 2380.02
   992.3 2381.78  1061.4  2380.4  1073.8 2383.14  1086.3 2392.02  1147.5 2399.43
#Mann= 5 ,-1,0
       0      .1       0   415.7    .045       0   462.4      .1       0
  864.19     .06       0  994.19      .1       0
Bank Sta=415.7,462.4
XS Rating Curve= 0 ,0
Exp/Cntr(USF)=0,0
Exp/Cntr=0.3,0.1

Type RM Length L Ch R = 1 ,38138   ,216.5,208.6,207.9
XS GIS Cut Line= 3
2363719.89717875710858.0795960162363895.87937742710565.148046484
2364255.43222523709810.478721642
#Sta/Elev= 30
       0 2404.88    16.1  2404.5      29 2401.48      85 2396.16   122.4 2398.73
   164.4 2397.43   201.7 2405.51     218 2407.25   346.1 2401.03   403.7 2410.07
   421.4 2415.41     426 2414.73     435 2405.71   452.5 2383.68     480 2377.07
   532.2 2377.33   638.6 2378.46     678 2375.41   696.2 2375.76     705 2381.53
   711.1 2382.91   770.2 2383.12   802.5 2380.42   829.1 2381.55   864.5 2378.93
   917.7 2378.52   974.8 2381.51  1049.2 2379.22  1112.7 2397.79  1177.7 2408.31
#Mann= 5 ,-1,0
       0      .1       0     480    .045       0   532.2      .1       0
  801.73     .06       0 1021.73      .1       0
Bank Sta=480,532.2
XS Rating Curve= 0 ,0
Exp/Cntr=0.3,0.1

Type RM Length L Ch R = 1 ,37929   ,609.2,615.8,603
XS GIS Cut Line= 3
2363918.98977604711086.6975468812364201.56325003710356.482925982
2364428.46065208709837.000120087
#Sta/Elev= 30
       0 2401.95   113.1 2399.02   250.4 2400.25     435  2393.9   486.3 2390.85
   499.2  2388.4   507.7 2377.85   512.3 2375.49   537.1  2375.4   602.3 2375.36
   619.3 2377.68     636 2377.82   700.7 2374.57   760.8 2374.85   778.3 2379.07
     791 2380.08   878.3 2377.65   939.4 2378.72   991.7 2376.06  1022.3 2378.15
  1074.7 2377.42  1099.3 2379.23  1144.5 2377.37  1166.3 2378.72  1188.2 2377.01
  1218.7 2380.28  1244.9 2379.54  1284.2 2392.59  1322.2 2408.93  1349.9 2415.33
#Mann= 10 ,-1,0
       0      .1       0      60     .06       0     160     .05       0
     270      .1       0     300     .05       0     380      .1       0
   537.1    .045       0   602.3      .1       0 1012.98     .06       0
 1122.98      .1       0
Bank Sta=537.1,602.3
XS Rating Curve= 0 ,0
Exp/Cntr(USF)=0,0
Exp/Cntr=0.3,0.1

Type RM Length L Ch R = 1 ,37313   ,198.7,210.6,215.4
XS GIS Cut Line= 4
2364159.59689251711425.2261642332364598.84476791710625.067614129
 2364688.3729973710350.8874116452364898.20478491710057.122908984
#Sta/Elev= 30
       0 2410.32    42.8 2396.53    56.4 2387.68    68.2 2386.21     105 2373.39
   115.4 2372.84   369.7 2372.51   492.9 2374.29   589.6 2372.93   781.1 2375.47
   862.5 2373.31   898.9 2370.31   925.3 2372.72   942.1 2371.23     959 2372.97
  1007.3 2370.69  1051.5 2370.08  1058.8 2370.67  1076.8 2374.23  1110.4 2374.91
  1139.9  2371.2  1180.2 2375.32  1190.4 2373.49  1205.2 2375.38    1223 2373.43
  1390.1 2374.25  1400.2 2378.94  1454.6 2415.15  1498.3  2438.5  1562.2 2477.76
#Mann= 9 ,-1,0
       0      .1       0     540     .06       0     670      .1       0
     750     .06       0     790      .1       0  1007.3    .045       0
  1058.8      .1       0 1102.79     .06       0 1251.22      .1       0
Bank Sta=1007.3,1058.8
XS Rating Curve= 0 ,0
Exp/Cntr(USF)=0,0
Exp/Cntr=0.3,0.1

Type RM Length L Ch R = 1 ,37103   ,137.1,132.6,135.7
XS GIS Cut Line= 3
2364213.68158753711444.5211456912364694.07723404710760.978898537
     2365071.166       710313.14
#Sta/Elev= 30
       0 2400.75    27.2 2393.12    48.1 2384.49    61.6 2383.39    73.9  2377.6
      97 2371.71   331.3 2370.75   352.2 2371.01   390.3 2374.02   421.7 2374.44
     493 2370.02   748.7 2374.53   776.5 2372.28     834  2371.9   844.9 2369.61
     868    2369   908.4 2372.35   938.1 2369.09   955.5 2368.76  1015.7 2369.18
  1039.1 2373.87  1122.8 2380.15  1154.2 2380.37  1180.6 2383.83  1198.9  2389.7
  1205.9 2390.55  1293.9 2394.63    1348 2394.57  1405.2 2398.34  1420.9 2400.75
#Mann= 9 ,-1,0
       0      .1       0      20     .08       0     140      .1       0
     500     .06       0     620      .1       0   938.1    .045       0
  1015.7      .1       0 1025.47     .06       0 1175.47      .1       0
Bank Sta=938.1,1015.7
XS Rating Curve= 0 ,0
Exp/Cntr=0.3,0.1

Type RM Length L Ch R = 1 ,36970   ,225.7,231.5,234.6
XS GIS Cut Line= 2
2364271.23346345711508.3252115732365019.03853504710571.320759969
#Sta/Elev= 30
       0 2411.83    31.4    2402    51.3 2393.84    70.6 2381.84    80.8 2380.51
    91.1 2374.42   106.4 2370.26     205 2369.92   234.3 2372.75   270.1 2371.01
   347.3 2371.99     367  2369.1   413.4 2368.79   597.7 2372.07   649.2 2370.77
   713.3 2372.32     741  2370.3   814.1 2371.51     828 2369.99   885.2 2372.45
   894.5 2372.19   904.7 2368.55   919.62367.605   942.2 2367.46   995.4 2367.73
    1066 2373.95  1142.9  2378.2  1147.1 2380.43  1169.9 2399.57  1198.8 2417.02
#Mann= 9 ,-1,0
       0      .1       0     110     .08       0     230      .1       0
     480     .06       0     610      .1       0   919.6    .045       0
   995.4      .1       0    1030     .06       0    1190      .1       0
Bank Sta=919.6,995.4
XS Rating Curve= 0 ,0
Exp/Cntr(USF)=0,0
Exp/Cntr=0.3,0.1

Type RM Length L Ch R = 1 ,36739   ,278.5,298.3,312.3
XS GIS Cut Line= 2
2364368.98228482711581.7901001442365169.58786813710783.544790257
#Sta/Elev= 30
       0 2406.87    23.5 2395.94    34.9 2392.85      44 2387.74    53.6  2384.7
    64.9 2377.71    76.2 2376.49    91.5 2371.22   148.2  2367.7   289.8  2367.2
   733.2 2371.87   771.3 2371.77     794 2369.03     801 2370.36   851.2 2368.21
     871 2369.08   882.3 2366.32   902.1 2369.48     913  2366.1   969.6 2365.57
   992.6 2366.57  1006.8  2368.8  1037.6 2367.17    1052 2372.32  1063.4 2373.78
  1066.2 2375.38  1077.7 2392.64  1083.4 2399.35  1108.6 2421.93  1130.6 2444.25
#Mann= 8 ,-1,0
       0      .1       0     210     .08       0     220      .1       0
     350     .06       0     490      .1       0     913    .045       0
   992.6      .1       0    1050     .06       0
Bank Sta=913,992.6
XS Rating Curve= 0 ,0
Exp/Cntr=0.3,0.1

Type RM Length L Ch R = 1 ,36440   ,187.5,189.6,191
XS GIS Cut Line= 5
2364516.66362381711693.8578296542364859.47049964 711394.72236751
2365093.28267323711190.7087469872365259.48912975711135.306594812
2365316.03525923711088.783092256
#Sta/Elev= 30
       0 2422.95    19.3 2414.01    61.9 2389.85    80.1 2370.77    85.2 2369.16
    94.9 2368.82   110.5 2364.32   142.7 2364.02   158.9 2366.51   195.7 2366.97
   376.3 2367.54   386.9 2366.67     433 2368.22   583.3 2367.59   615.3 2368.88
   662.9 2367.58   753.2 2369.58   770.1  2366.6   814.7 2365.58   827.4 2363.64
   856.9 2363.31   881.3 2364.22   895.3 2363.96     899 2364.96   907.5 2370.74
   915.9 2370.67   921.9 2372.06   926.9 2375.16   951.7 2396.24  1013.7 2428.78
#Mann= 9 ,-1,0
       0      .1       0     110     .08       0     140      .1       0
     270     .06       0     410      .1       0  785.28     .06       0
   827.4    .045       0   881.3     .06       0  885.28      .1       0
Bank Sta=827.4,881.3
XS Rating Curve= 0 ,0
Exp/Cntr(USF)=0,0
Exp/Cntr=0.3,0.1

Type RM Length L Ch R = 1 ,36251   ,397.7,394.7,393
XS GIS Cut Line= 4
2364630.51585311711798.7897533972364906.16052839711577.462803416
2365142.22124098711367.7647916472365420.64530622711291.989086636
#Sta/Elev= 30
       0 2454.45    21.7 2440.57    32.9 2431.43    66.5 2407.85    79.1 2387.77
   101.9 2372.02   110.4 2367.04   117.6 2364.75   130.4 2364.62   147.4 2361.94
   198.6 2365.19   264.5 2364.41     399 2367.09   546.7 2367.68   588.8 2366.34
   607.7 2368.01   650.5  2364.2   661.2 2361.06   671.3 2364.06   683.7 2364.82
   731.6 2362.33   796.8 2362.24   803.9 2363.24   813.1 2369.26   829.4 2370.74
   857.8 2397.18     891 2414.92   922.8 2428.17   936.6 2430.44   957.8 2437.82
#Mann= 7 ,-1,0
       0      .1       0   363.5     .06       0   493.5      .1       0
   731.6    .045       0   796.8      .1       0  809.25     .06       0
  839.25      .1       0
Bank Sta=731.6,796.8
XS Rating Curve= 0 ,0
Exp/Cntr=0.3,0.1

Type RM Length L Ch R = 1 ,35856   ,260.4,259.6,260.2
XS GIS Cut Line= 2
2364715.76599129711969.3853612522365654.56895217711571.482119553
#Sta/Elev= 30
       0 2462.95   135.1 2437.29   182.9 2425.71   192.7 2421.31   213.3 2405.31
   230.7 2394.08   259.8 2376.98   282.8 2365.79   293.4 2363.38   338.8 2362.61
   369.5 2358.78     400 2359.68   417.5 2363.18     461 2364.08   495.7  2362.2
   526.1 2364.25   565.2 2363.71   573.9 2362.89   583.3 2359.79   641.2 2359.94
   711.4 2361.31   731.8 2359.47   747.7 2359.86   763.3 2367.75   775.5 2369.75
   790.7 2381.31   838.9  2404.7     860 2412.65   977.9 2461.81  1019.6 2477.78
#Mann= 4 ,-1,0
       0      .1       0   583.3    .045       0   641.2     .06       0
     860      .1       0
Bank Sta=583.3,641.2
XS Rating Curve= 0 ,0
Exp/Cntr(USF)=0,0
Exp/Cntr=0.3,0.1

Type RM Length L Ch R = 1 ,35597   ,240.1,249.1,253.9
XS GIS Cut Line= 3
     2365029.716      712103.3172365348.73385605711932.873953197
2365727.70747512711784.818906394
#Sta/Elev= 30
       0 2420.93    47.7 2417.59    61.7  2413.6    79.9 2403.34   102.6 2384.05
   115.7 2370.89   130.5 2360.41   134.3 2358.21   152.4 2356.59   168.9    2360
   216.7 2357.21   274.9 2359.79   284.2 2357.91   320.2 2357.42   337.4  2357.9
   349.2 2360.36   373.4 2360.36   382.6 2357.84   395.5 2360.47   425.5 2361.17
   455.6  2360.9     474 2357.72   523.3 2357.38   532.9 2358.05   541.5 2366.79
   558.6 2370.38   571.5 2382.37   614.2 2405.61   691.8 2433.95   768.6 2474.22
#Mann= 5 ,-1,0
       0      .1       0  421.69     .06       0     474    .045       0
   523.3     .06       0  631.69      .1       0
Bank Sta=474,523.3
XS Rating Curve= 0 ,0
Exp/Cntr=0.3,0.1

Type RM Length L Ch R = 1 ,35347   ,177.9,184,188.1
XS GIS Cut Line= 2
2365052.36424312712165.3226064292365816.08670742712100.079983851
#Sta/Elev= 30
       0 2415.09    15.9 2413.79      60 2403.68    72.1 2397.17    96.2 2386.82
   120.2 2365.24   124.3 2360.61   128.3 2358.79   140.3 2358.12   152.4 2355.03
   164.4 2357.25   192.3 2359.45   224.6 2360.06   236.7 2359.16   244.7 2356.13
   260.8 2355.41   373.2 2358.44   421.3 2358.12     443 2356.11   484.5 2355.72
   501.6 2360.13   509.7 2365.71   525.7 2368.22   537.8  2381.2   553.8 2394.92
   569.9 2405.25     598 2425.49   646.2 2447.08   690.3 2468.52   766.5 2513.26
#Mann= 4 ,-1,0
       0      .1       0     443    .045       0   484.5     .06       0
     650      .1       0
Bank Sta=443,484.5
XS Rating Curve= 0 ,0
Exp/Cntr(USF)=0,0
Exp/Cntr=0.3,0.1

Type RM Length L Ch R = 1 ,35163   ,234.5,247,249.3
XS GIS Cut Line= 3
2364986.60823756712236.4311427732365358.13214159712285.446094788
2365760.24185545712350.743475712
#Sta/Elev= 30
       0  2412.5      27 2408.74    58.1 2401.41    66.9 2400.71    98.4  2391.1
   126.4 2378.57   138.8 2375.63   155.3    2364     163  2360.5   187.4 2357.74
   226.6 2357.67   235.6 2354.33   251.6 2353.82   292.1 2353.97   384.9 2357.12
   425.4 2354.01   461.9 2356.19   484.4 2354.52   522.7 2354.34     547  2357.4
   555.1 2363.43   571.1 2366.51   575.4 2368.46   587.5 2379.14     620 2401.27
   660.5 2432.25   679.6 2444.61     701 2461.09   750.1 2491.92   782.1 2513.65
#Mann= 5 ,-1,0
       0      .1       0   484.4    .045       0   522.7      .1       0
  524.74     .06       0  624.74      .1       0
Bank Sta=484.4,522.7
XS Rating Curve= 0 ,0
Exp/Cntr=0.3,0.1

Type RM Length L Ch R = 1 ,34916   ,209.3,215.6,219.3
XS GIS Cut Line= 2
2364971.77041523 712307.321255572365658.73685296712664.236779085
#Sta/Elev= 30
       0 2398.25    28.4 2390.98    52.1 2386.87    84.7 2376.98    99.6 2375.56
   113.1  2371.1   144.1  2357.4   161.9 2354.01   194.5 2356.06   225.8 2353.05
   283.5 2352.42   311.5 2355.73     325 2353.84   352.1 2355.41   374.6  2353.5
   397.1 2355.73   419.7 2355.88   455.2 2352.88   514.3 2352.51   523.3 2353.98
   532.4 2362.16   550.4 2364.49   553.4 2366.38     600  2408.3   651.3 2454.83
   672.1 2470.77   690.1 2486.91   730.7 2513.78   750.2 2531.11   774.2 2555.02
#Mann= 5 ,-1,0
       0      .1       0   455.2    .045       0   514.3      .1       0
     600     .06       0     660      .1       0
Bank Sta=455.2,514.3
XS Rating Curve= 0 ,0
Exp/Cntr(USF)=0,0
Exp/Cntr=0.3,0.1

Type RM Length L Ch R = 1 ,34701   ,334.7,339.8,341.5
XS GIS Cut Line= 3
2364892.22447571 712380.916237562365461.93290639712848.035000591
2365584.62138033  712935.2135705
#Sta/Elev= 30
       0  2385.9    82.4 2372.51   116.7 2372.72   150.8 2367.57   187.7 2351.49
   258.6 2354.08     273 2351.36   310.3 2355.39   347.4 2354.93   366.3 2351.52
   434.4 2350.31     472 2354.14   517.7 2351.95   568.2 2350.79   574.5 2352.81
   582.8 2360.56   594.2 2361.92   599.9 2365.84   614.1 2381.13   636.2 2398.69
   667.2 2426.86   685.1 2451.25   698.2 2464.61   756.4 2512.57   770.7 2529.62
   799.4 2552.08     808 2563.62   813.1    2568   833.8 2577.57   887.2 2596.62
#Mann= 4 ,-1,0
       0      .1       0   517.7    .045       0   568.2     .06       0
     680      .1       0
Bank Sta=517.7,568.2
XS Rating Curve= 0 ,0
Exp/Cntr=0.3,0.1

Type RM Length L Ch R = 1 ,34361   ,214.1,221.4,224
XS GIS Cut Line= 2
2364733.82673289712514.5625272882365248.09211086713174.664355724
#Sta/Elev= 30
       0  2392.6    23.6 2385.13    64.2 2375.63   114.7 2357.03   140.2 2351.34
   153.5 2353.57   165.6 2350.73   185.9 2352.15   211.6 2349.18   237.3 2349.21
   251.8 2350.01     267 2353.18   285.7  2348.9   307.6 2352.79   342.3 2352.88
   444.5 2348.34   490.9 2347.98   525.1 2348.43   537.5 2348.51   550.9 2353.55
   571.2 2354.18   576.6 2356.33     622 2392.84     627 2399.55   642.2 2424.32
   656.2 2441.48   696.1 2474.44   778.3  2525.8   815.8 2542.27   836.8 2546.14
#Mann= 4 ,-1,0
       0      .1       0   444.5    .045       0   525.1     .06       0
     630      .1       0
Bank Sta=444.5,525.1
XS Rating Curve= 0 ,0
Exp/Cntr(USF)=0,0
Exp/Cntr=0.3,0.1

Type RM Length L Ch R = 1 ,34140   ,231.1,218.2,221
XS GIS Cut Line= 4
2364559.67085495712592.3198947922364770.37714647712888.321839446
2364939.16637873   713163.1213282365028.82487005713308.690446146
#Sta/Elev= 30
       0 2421.94    69.8 2393.94     125 2375.51   145.7 2364.59   159.5 2360.39
   170.2  2353.6   181.7 2352.05   192.5 2347.53   228.5 2349.14   247.6 2347.42
   269.9 2350.11   304.4 2347.54   334.9 2352.17     369 2351.24   387.8 2346.76
   403.1 2348.56   430.1 2345.69   461.2 2347.24   525.2 2347.17   557.2 2350.73
   577.6 2347.08   594.4 2348.36   613.1 2363.53   627.2 2385.16     659 2410.79
     754 2470.29   796.3 2485.75   817.4 2491.08   833.9 2493.51   856.8 2493.13
#Mann= 5 ,-1,0
       0      .1       0  443.34     .06       0   461.2    .045       0
   525.2     .06       0  623.34      .1       0
Bank Sta=461.2,525.2
XS Rating Curve= 0 ,0
Exp/Cntr=0.3,0.1

Type RM Length L Ch R = 1 ,33921   ,548.1,557.3,546.8
XS GIS Cut Line= 4
2364365.49672645712822.3508110722364560.28225339712990.813969508
2364709.00248107 713146.25278129 2364949.4671917713381.210666481
#Sta/Elev= 30
       0 2417.93    89.9 2384.74   125.8  2363.7   159.9 2347.58   179.7 2345.41
   193.9 2347.97   205.2 2347.78   236.7 2345.09   263.2 2349.17   290.2 2349.52
   310.6 2345.44     321 2345.18   343.8 2344.03   380.8 2344.66   399.2 2347.06
   414.7 2345.05   442.5 2345.14     460 2348.45   502.4 2345.76   536.4  2351.4
     542 2354.34   561.8 2372.14   581.6 2383.73   616.9 2403.61   628.1 2407.21
     658 2421.84   717.4 2443.29   756.7 2451.48   774.5 2457.68   808.9 2463.98
#Mann= 5 ,-1,0
       0      .1       0     321    .045       0   380.8      .1       0
  482.65     .06       0  622.65      .1       0
Bank Sta=321,380.8
XS Rating Curve= 0 ,0
Exp/Cntr(USF)=0,0
Exp/Cntr=0.3,0.1

Type RM Length L Ch R = 1 ,33364   ,262.4,247.2,231.9
XS GIS Cut Line= 3
2363991.71909367713201.3929175532364448.92043689 713518.21051652
2364770.45060372 713508.34812977
#Sta/Elev= 30
       0 2490.35    62.8 2454.43   112.5 2420.16     141 2395.18   161.1 2380.75
   195.2 2348.94   214.7 2341.55   224.4 2340.56   267.5 2340.45   287.6    2344
   308.6 2339.74   329.7 2341.38   341.2 2344.58   355.8 2345.33   404.5 2344.98
   422.7 2342.98   443.4 2345.98   517.6 2344.76   540.6 2346.94   715.6 2346.28
   731.6 2344.41   743.6 2344.73   755.6 2342.93   775.6 2343.04   779.6 2344.06
   787.6 2349.06   803.6 2351.68   815.6 2360.67   839.3 2371.35   877.9    2386
#Mann= 5 ,-1,0
       0      .1       0   224.4    .045       0   267.5      .1       0
  726.24     .06       0  826.24      .1       0
Bank Sta=224.4,267.5
XS Rating Curve= 0 ,0
Exp/Cntr(USF)=0,0
Exp/Cntr=0.3,0.1

Type RM Length L Ch R = 1 ,33117   ,237.8,236.7,235.7
XS GIS Cut Line= 3
2363854.52408096713562.6130847812364364.13446248713575.582190758
2364856.19456845713662.783809242
#Sta/Elev= 30
       0  2513.5     9.7 2506.48    17.7 2497.23    44.2 2477.59   100.9 2439.18
   125.7 2417.84   149.7 2393.38   181.7 2368.33   193.7 2356.18   201.7 2344.93
   205.7 2341.32   209.7 2338.88   226.5 2339.06   277.3 2337.66   286.5 2337.89
   313.8 2344.25   361.8 2342.47   402.1 2343.21   453.8 2340.33   497.8 2344.86
   552.6 2345.38   757.6 2344.91   769.8 2341.14   777.9 2340.78   798.2 2343.04
   822.6 2342.88   842.9  2347.9   859.2 2348.68   873.2 2356.52  1009.5 2404.71
#Mann= 5 ,-1,0
       0      .1       0   226.5    .045       0   286.5      .1       0
  769.78     .06       0  869.78      .1       0
Bank Sta=226.5,286.5
XS Rating Curve= 0 ,0
Exp/Cntr=0.3,0.1

Type RM Length L Ch R = 1 ,32880   ,248.5,241.6,238.9
XS GIS Cut Line= 2
2363912.75198815713806.8073931812364865.62172806 713801.54291948
#Sta/Elev= 30
       0 2459.51      30 2440.69    50.1 2426.07   111.4 2376.41   147.4 2338.36
   151.4 2336.81   159.4 2336.61   191.4 2336.26   231.4 2336.28   243.4 2336.98
   251.4 2340.59   259.4 2341.53   303.4 2340.56   335.4 2337.08   363.4 2336.98
   383.4 2341.54   420.1 2340.48   459.4 2343.55   499.4 2342.18   579.4    2342
   651.4 2343.22   747.4 2338.68     762 2341.61   787.4 2342.05   799.4 2346.26
   815.4 2346.53   851.4 2360.51   879.4 2374.15   931.4 2388.77   952.9 2391.89
#Mann= 7 ,-1,0
       0      .1       0   159.4    .045       0   231.4      .1       0
     510     .12       0     610      .1       0     710     .06       0
     810      .1       0
#XS Ineff= 1 ,-1
  483.16  636.99 2352.08
Permanent Ineff=
       F
Bank Sta=159.4,231.4
XS Rating Curve= 0 ,0
Exp/Cntr(USF)=0,0
Exp/Cntr=0.3,0.1

Type RM Length L Ch R = 1 ,32639   ,257.1,252.1,249.8
XS GIS Cut Line= 3
 2363937.5153353714076.2097456562364451.88473801714001.015745656
2364952.43905594713891.280533703
#Sta/Elev= 30
       0 2467.11     6.7 2463.19    14.8 2453.28    43.1 2426.39     132 2363.16
   163.7 2336.59   176.5 2334.16   212.6 2333.97   233.1    2334   249.3  2334.4
   261.4 2338.48     322 2338.54   338.2  2334.9   366.5 2339.47   427.2 2336.67
   471.6 2337.46   484.7 2335.24     504  2340.2   548.8 2340.81   593.9 2340.84
   630.7 2337.47   683.9 2340.86   712.6 2336.94   778.6 2337.86   823.2 2345.86
   839.5 2358.97   868.2 2374.57   917.3 2388.06   974.7  2397.4  1032.3 2402.39
#Mann= 7 ,-1,0
       0      .1       0   176.5    .045       0   233.1      .1       0
  589.84     .12       0  689.84      .1       0  789.84     .06       0
  889.84      .1       0
Bank Sta=176.5,233.1
XS Rating Curve= 0 ,0
Exp/Cntr=0.3,0.1

Type RM Length L Ch R = 1 ,32387   ,263.4,258.1,254.2
XS GIS Cut Line= 2
2364002.24804107714349.0481843972364913.00199137714091.088973042
#Sta/Elev= 30
       0 2452.89    43.6 2425.69      56 2413.35    85.7 2388.45   114.3 2371.05
   124.8 2362.29   143.4 2354.18   168.3 2332.78   189.1  2332.3   190.3 2332.27
   246.6 2332.51   268.1 2336.12   301.3 2336.19   318.9 2332.86   338.7 2336.67
   376.2 2339.73   432.2  2340.2   496.7 2338.37   650.5 2338.95   712.9  2336.1
   725.4 2333.66   746.2 2334.47   762.8 2336.81   775.3 2341.01   796.1 2341.31
   816.8 2352.38   841.8 2358.97   879.4 2376.98   911.8 2386.99   946.6 2393.05
#Mann= 5 ,-1,0
       0      .1       0   189.1    .045       0   246.6      .1       0
     740     .06       0     850      .1       0
Bank Sta=189.1,246.6
XS Rating Curve= 0 ,0
Exp/Cntr(USF)=0,0
Exp/Cntr=0.3,0.1

Type RM Length L Ch R = 1 ,32129   ,284.8,278.8,273.5
XS GIS Cut Line= 3
2364097.35223992714624.1033323482364513.66571623714436.749665878
2364987.09685959714203.307760666
#Sta/Elev= 30
       0  2475.4     7.5 2471.14    29.4 2452.98    42.6 2444.92   139.1 2372.17
   164.7 2346.16   174.2 2333.83   178.6 2331.64   188.9 2330.29   253.1 2329.76
   257.5 2329.85   275.1 2333.64   292.6 2331.98   314.5 2335.23   393.5 2335.78
   436.9 2332.32     467 2336.61   523.8 2337.78   646.3 2336.52   682.3 2332.27
   704.6 2334.55   731.4 2334.44   749.2 2337.76   793.8 2338.45   798.6 2339.04
   807.2 2342.71   838.4 2358.62   874.1 2379.47   887.5 2385.13   984.4 2394.53
#Mann= 5 ,-1,0
       0      .1       0   188.9    .045       0   257.5      .1       0
  686.53     .06       0  796.53      .1       0
Bank Sta=188.9,257.5
XS Rating Curve= 0 ,0
Exp/Cntr=0.3,0.1

Type RM Length L Ch R = 1 ,31850   ,266.7,260.3,255.9
XS GIS Cut Line= 2
2364260.82734478714894.3877260642365108.37990132714325.575716197
#Sta/Elev= 30
       0 2476.88   127.2 2383.01   174.4 2331.83   182.3 2328.56   193.5 2328.57
   201.5 2327.82   254.1 2327.91   273.8 2331.64   296.5 2329.31   341.2 2333.25
   372.3 2332.52   395.3 2334.73   456.9 2334.41   481.8 2332.81   510.6 2335.31
   542.3 2333.73   577.3 2335.52   631.7 2335.61   646.1 2334.35   659.2 2329.99
   673.6 2329.84   688.1 2332.82   726.6 2337.03   750.7 2350.38     770  2357.5
   784.2  2360.6   842.1 2380.07   885.1 2389.71   978.4 2398.24  1020.7 2404.17
#Mann= 5 ,-1,0
       0      .1       0   193.5    .045       0   254.1      .1       0
     670     .06       0     750      .1       0
Bank Sta=193.5,254.1
XS Rating Curve= 0 ,0
Exp/Cntr(USF)=0,0
Exp/Cntr=0.3,0.1

Type RM Length L Ch R = 1 ,31589   ,200,201.1,201.9
XS GIS Cut Line= 3
2364386.01133412  715173.05257052364527.78261848715050.198763031
2365223.52147926714389.544236379
#Sta/Elev= 30
       0 2519.57    18.5  2507.8    52.5 2481.29     112 2439.58   200.7 2370.65
   215.7 2356.49   245.2 2337.05   264.6 2327.26   270.4 2326.67   322.7 2326.27
   348.1 2327.21   370.2 2330.29   403.6 2330.91   447.4 2328.93   469.5 2332.67
   508.1 2333.66   585.3 2331.02   686.6 2334.79   756.3 2329.91   772.8 2334.26
   788.4 2335.33   799.7 2343.11   816.7 2350.65   881.8  2372.3   966.7 2390.29
   993.5 2398.42  1065.7  2412.1  1089.5 2414.07  1114.8 2412.37    1147 2417.95
#Mann= 5 ,-1,0
       0      .1       0   270.4    .045       0   348.1      .1       0
   737.6     .06       0   877.6      .1       0
Bank Sta=270.4,348.1
XS Rating Curve= 0 ,0
Exp/Cntr=0.3,0.1

Type RM Length L Ch R = 1 ,31388   ,221.9,213.6,216.5
XS GIS Cut Line= 4
2364519.17224169 715336.293470782364912.58913349714958.464889864
2365031.83318287714956.2566667282365265.38411131 714748.14056759
#Sta/Elev= 30
       0 2520.42      34 2495.44    67.9 2473.02   101.2 2448.14   114.2 2435.61
   138.7 2416.43   173.3  2383.7   212.3 2350.85   239.9 2332.51   246.2 2329.93
   288.6 2325.66   328.6 2325.29   396.1 2326.11   404.6 2328.58   438.6 2328.01
   469.7 2330.69   500.5 2329.31   528.3 2331.84   549.1 2331.95   565.1 2329.59
   609.2 2326.94   649.1 2331.12   814.5 2330.64   861.8 2332.55     874 2337.41
     891  2349.4   933.9 2368.45   949.1 2376.75   959.9 2377.88   977.6 2384.73
#Mann= 5 ,-1,0
       0      .1       0   288.6    .045       0   396.1      .1       0
  774.73     .06       0  904.73      .1       0
#XS Ineff= 2 , 0
                          652.48         2342.07
Permanent Ineff=
       F       F
Bank Sta=288.6,396.1
XS Rating Curve= 0 ,0
Exp/Cntr(USF)=0,0
Exp/Cntr=0.3,0.1

Type RM Length L Ch R = 1 ,31175   ,252,262,267.9
XS GIS Cut Line= 3
2364625.80319017715518.8249520152365161.47028732715015.135664696
2365457.98571564714772.096522515
#Sta/Elev= 30
       0 2543.42    14.2  2538.8    53.8 2513.74    84.2 2492.62     124 2458.94
   130.9 2455.57     157 2436.14   183.9 2412.31   211.9 2378.24   222.9 2362.44
   251.9  2339.4   268.8 2328.97     300 2323.58   311.9 2326.21   359.4 2327.64
   409.6 2324.18   495.2  2323.9   519.4    2324   530.4 2327.34   629.2 2330.74
   701.8 2329.73   781.2 2331.27   847.4 2329.17   889.8 2331.07   902.4 2334.63
   921.4 2347.26   950.8 2362.24  1011.5 2379.79  1066.5 2399.61  1118.7 2415.57
#Mann= 5 ,-1,0
       0      .1       0   409.6    .045       0   495.2      .1       0
  795.28     .06       0  925.28      .1       0
#XS Ineff= 2 , 0
                          826.91         2367.53
Permanent Ineff=
       F       F
Bank Sta=409.6,495.2
XS Rating Curve= 0 ,0
Exp/Cntr=0.3,0.1

Type RM Length L Ch R = 1 ,30913   ,208,195.8,193.1
XS GIS Cut Line= 3
2364783.21573502715555.5517813542364912.01291918715542.117885117
2365589.32501129 715090.31914063
#Sta/Elev= 30
       0 2456.65    45.2 2422.81    86.8 2382.68   106.2 2357.35   144.1 2328.19
   158.5 2323.46   211.4 2321.16   230.7 2324.42   249.9  2322.4   291.8 2326.78
   307.6 2325.55   320.7 2321.85   347.4 2324.81   361.9 2322.56   455.6  2322.1
   467.8  2322.4   499.9 2327.92   539.9 2325.09   557.6 2326.52   591.3 2325.69
   606.9 2328.97   655.2 2328.92   681.2 2325.37   715.8 2326.26   738.9 2329.25
   764.8 2346.58   778.8 2351.82   888.9 2372.42   916.9 2380.39   943.7 2390.67
#Mann= 5 ,-1,0
       0      .1       0   361.9    .045       0   455.6      .1       0
   719.5     .06       0   839.5      .1       0
#XS Ineff= 2 , 0
                          655.74         2349.55
Permanent Ineff=
       F       F
Bank Sta=361.9,455.6
XS Rating Curve= 0 ,0
Exp/Cntr(USF)=0,0
Exp/Cntr=0.3,0.1

Type RM Length L Ch R = 1 ,30717   ,330.9,358.2,386.8
XS GIS Cut Line= 3
2364866.22305848715695.5106460462365231.46836622715564.990347822
     2365637.826      715223.219
#Sta/Elev= 30
       0 2403.64    19.1 2392.74    27.6 2389.49      53 2372.44    57.3 2368.11
      70 2349.13    95.5 2328.82   112.5 2320.65   125.3  2319.3   176.2 2319.44
   197.5 2322.65   231.4 2321.49   269.7 2323.66   297.5 2319.09   320.7 2323.49
     400 2324.58   414.9 2323.43   436.5 2324.69   453.5 2321.88   529.9 2321.69
   540.4 2321.26   564.2 2324.91   648.6 2322.97   707.6 2328.25   766.6 2327.01
   811.2 2339.45     854 2347.02   869.6 2351.22   903.4 2364.63   918.8 2372.51
#Mann= 5 ,-1,0
       0      .1       0   453.5    .045       0   529.9      .1       0
  617.87     .06       0  747.87      .1       0
#XS Ineff= 2 , 0
                          691.92         2346.43
Permanent Ineff=
       F       F
Bank Sta=453.5,529.9
XS Rating Curve= 0 ,0
Exp/Cntr=0.3,0.1

Type RM Length L Ch R = 1 ,30359   ,149.6,160.1,171.9
XS GIS Cut Line= 4
2364857.86145058715739.8850430092365216.82488629715770.478517644
2365590.06527682715829.6259019362365861.90655431715844.903210384
#Sta/Elev= 30
       0 2401.04    50.5 2374.38    70.6 2358.56    78.6 2354.45   102.7 2333.46
   126.8 2318.23     187 2322.94   207.1  2320.1   239.2 2322.25   287.4 2321.52
   303.4 2317.06   315.5 2319.86   347.6 2322.07     397 2320.65   416.3 2321.84
   432.5  2318.2   449.5 2321.25   480.9 2322.86   497.3  2318.4   521.6 2320.68
   536.9 2319.65   596.9  2319.7   618.8 2327.49   695.7 2333.09   760.3 2332.72
   792.8 2347.58   828.4 2352.07   920.6 2356.62   963.5 2351.98  1010.4 2353.51
#Mann= 6 ,-1,0
       0      .1       0   536.9    .045       0   596.9      .1       0
  650.26     .06       0  748.16      .1       0  848.16     .06       0
Bank Sta=536.9,596.9
XS Rating Curve= 0 ,0
Exp/Cntr(USF)=0,0
Exp/Cntr=0.3,0.1

Type RM Length L Ch R = 1 ,30199   ,214.7,224.5,225.3
XS GIS Cut Line= 3
2364813.69362922715823.9872185932365216.50098008715855.887364141
2365779.56846375716224.921384063
#Sta/Elev= 30
       0 2405.32    34.6 2396.92   102.8 2370.55   118.9 2362.04   138.9  2347.7
     151  2340.7     171 2324.33   195.1 2316.33   219.2 2318.78   243.2 2316.86
   256.2 2319.79   283.4  2320.6   395.7 2321.06   416.3 2318.25   450.2 2321.77
   489.8 2317.98   561.5  2317.9   581.6 2326.03   644.6 2327.18     659 2329.06
   720.2 2328.17   762.4  2333.1   800.5 2330.15   812.1 2333.66   862.8 2337.87
     888 2347.91   916.1 2353.38   948.9 2362.17  1015.8 2391.99  1077.3 2424.31
#Mann= 5 ,-1,0
       0      .1       0   489.8    .045       0   561.5      .1       0
  594.07     .06       0  754.07      .1       0
Bank Sta=489.8,561.5
XS Rating Curve= 0 ,0
Exp/Cntr=0.3,0.1

Type RM Length L Ch R = 1 ,29974   ,228.1,190.7,169
XS GIS Cut Line= 4
2364793.68421182715873.3589975212364980.42900793715893.805508045
2365203.97752299716107.8123181932365521.57998646716159.610144852
#Sta/Elev= 30
       0 2405.34    54.8 2393.37   111.2 2376.14   132.7 2366.04   155.4 2352.59
   175.5 2338.56   187.6 2326.78     193 2322.78   209.9 2317.24   215.2 2315.95
   226.3 2315.82   244.8 2320.01   274.9 2317.56   331.6 2319.34   348.1 2318.55
     357 2315.87   370.2 2315.71   435.7 2316.62   447.8 2319.71   469.9 2319.79
     482 2322.77     534 2319.99   647.5 2322.26   720.4 2326.56   736.7 2326.06
   744.8    2328   756.6 2328.91   785.3 2327.15   801.9 2329.68   819.1 2330.45
#Mann= 4 ,-1,0
       0      .1       0     357    .045       0   435.7     .06       0
  707.33      .1       0
Bank Sta=357,435.7
XS Rating Curve= 0 ,0
Exp/Cntr(USF)=0,0
Exp/Cntr=0.3,0.1

Type RM Length L Ch R = 1 ,29783   ,100,93.8,91.7
XS GIS Cut Line= 4
2364872.65515941716223.849379799 2365113.8728936716117.327988107
2365233.69983898716162.8665481292365489.25685783716253.916449785
#Sta/Elev= 30
       0 2363.86    12.6 2362.65    25.9 2360.18    38.8 2356.65    47.6 2355.47
    56.3 2352.48    86.9 2333.17    95.7 2323.69     100 2317.46   105.6 2314.81
   126.3 2313.75   166.1 2313.84   200.6 2318.21   257.5 2320.67   274.7  2320.6
   293.3 2323.02   321.8 2322.26   327.4 2321.54   336.7 2318.79   342.1  2318.3
   360.3 2320.39   428.5 2319.09     454 2320.33   517.6 2321.32   550.5 2322.59
   572.9 2325.86   585.6 2325.51   594.1  2324.4   611.1 2325.28   663.2 2325.18
#Mann= 5 ,-1,0
       0      .1       0      50     .06       0   105.6    .045       0
   166.1     .06       0  373.69      .1       0
Bank Sta=105.6,166.1
XS Rating Curve= 0 ,0
Exp/Cntr(USF)=0,0
Exp/Cntr=0.3,0.1

Type RM Length L Ch R = 1 ,29690   ,80.7,119.1,142
XS GIS Cut Line= 4
2364927.28593454 716299.163421142365047.22687192 716232.05784232
2365141.27489072716177.3304539732365609.06765048716289.834504294
#Sta/Elev= 30
       0 2323.35    10.2 2323.61    19.4 2322.46    33.1  2315.4    37.7 2314.28
    46.9  2313.8     105 2313.92   115.6 2314.31   129.4  2319.1   146.1 2322.94
     167 2324.04   206.8 2322.39   231.1 2319.79   335.6 2320.05     348 2317.98
   376.8 2319.71   401.1 2319.26   454.1 2320.68   512.5 2324.97   530.4 2323.78
   590.7 2325.12   615.4 2324.31   619.5  2324.8   626.6    2328   644.2 2340.02
   652.4 2344.67   669.7 2361.04   681.2 2369.37   696.2 2375.28   727.4 2381.99
#Mann= 4 ,-1,0
       0      .1       0    37.7    .045       0     105     .06       0
  207.44      .1       0
Bank Sta=37.7,105
XS Rating Curve= 0 ,0
Exp/Cntr(USF)=0,0
Exp/Cntr=0.3,0.1

Type RM Length L Ch R = 1 ,29570   ,433.5,436,423.6
XS GIS Cut Line= 5
2364683.79039567716255.3508348692364866.09125878716310.878379013
2364950.04304769716359.4491395632365029.10924007716393.175461362
2365369.56120051716612.511205416
#Sta/Elev= 30
       0 2363.08    12.9  2357.5    21.3 2356.72    42.2 2362.52    58.9 2364.69
     114 2366.37   134.2 2362.62   159.3 2352.54   163.5 2349.62   180.2 2331.54
   197.6 2323.56   243.8 2322.15     264 2315.23   290.5 2313.85   360.6 2313.82
   432.6 2312.48   462.8 2313.43   477.1 2316.03   615.1 2315.14   624.6 2316.75
   653.1 2315.43   662.2 2311.98   667.4 2311.61   682.5 2311.82   699.9 2316.45
   705.5 2321.51   710.2 2327.72   720.7 2334.44   757.7    2368   778.5 2384.63
#Mann= 5 ,-1,0
       0      .1       0     140     .06       0  250.57      .1       0
   290.5    .045       0   360.6      .1       0
Bank Sta=290.5,360.6
XS Rating Curve= 0 ,0
Exp/Cntr(USF)=0,0
Exp/Cntr=0.3,0.1

Type RM Length L Ch R = 1 ,29134   ,185.8,194.7,204.8
XS GIS Cut Line= 2
2364548.17930018716458.9394991132365304.77640142716782.524929205
#Sta/Elev= 30
       0 2361.11    26.1 2354.85    43.5 2352.83    78.3 2342.67   117.5  2347.2
   156.6 2345.31   181.5 2337.51   202.8 2317.88   230.6 2319.19   251.6 2313.64
   303.4 2315.84   321.9 2313.65   417.6 2313.67   430.7 2311.45   439.4  2313.8
   452.4 2314.16     509 2310.11   535.1 2312.59   604.7    2313   617.8  2310.9
   646.5 2309.78   677.1 2311.06   696.1 2322.12   707.6 2333.28   720.8 2351.87
   727.9 2357.84   735.2 2369.91   739.1 2374.33   796.1 2410.99   822.9 2430.82
#Mann= 5 ,-1,0
       0      .1       0     180     .06       0     290      .1       0
   617.8    .045       0   677.1      .1       0
Bank Sta=617.8,677.1
XS Rating Curve= 0 ,0
Exp/Cntr=0.3,0.1

Type RM Length L Ch R = 1 ,28940   ,513.4,509.8,496.8
XS GIS Cut Line= 3
 2364574.1094754716582.1412089582364927.18719759716789.382480676
2365191.99548923716981.272547082
#Sta/Elev= 30
       0 2355.42       6 2354.39    62.2 2336.29    67.3 2333.55    76.8 2324.96
    97.3  2323.2   108.9 2315.86   111.9 2315.26     123 2316.45   146.2 2316.05
     174 2310.67   190.8 2312.64   255.5 2313.78   284.3 2312.49   353.7 2312.81
   373.4 2309.14   450.1 2308.31   486.5 2309.17   499.5 2308.05   521.7 2308.27
   530.3 2310.46     544 2311.64   548.9  2313.5   553.9 2317.94   561.8 2329.37
   573.2 2338.14   673.5 2403.01   687.8 2415.66   702.1 2425.33   736.4 2445.64
#Mann= 5 ,-1,0
       0      .1       0      50     .06       0     280      .1       0
   486.5    .045       0   521.7      .1       0
#XS Ineff= 2 , 0
          127.08 2335.38
Permanent Ineff=
       F       F
Bank Sta=486.5,521.7
XS Rating Curve= 0 ,0
Exp/Cntr(USF)=0,0
Exp/Cntr=0.3,0.1

Type RM Length L Ch R = 1 ,28430   ,192.6,191,190.1
XS GIS Cut Line= 2
 2364344.3327577717064.6464424272365046.01365155717219.666522951
#Sta/Elev= 30
       0 2328.93    69.5 2326.01      90 2317.62   110.4 2318.38     135 2315.08
   154.7 2314.43   168.1 2315.61   218.4 2311.16   235.2 2305.06   274.3 2305.17
   290.7 2306.86   298.9 2305.25   352.6 2305.58   372.6 2307.58   393.1 2305.88
   406.3 2308.52   483.2 2308.95   496.9 2306.67     516 2308.05   556.5 2307.41
   569.2 2304.48   593.8 2304.75   597.9 2305.98   632.9 2334.21     643 2340.82
   655.3 2351.05   663.5 2355.38   679.8 2370.16   708.3 2390.35   718.6 2400.24
#Mann= 7 ,-1,0
       0      .1       0      80     .06       0     180      .1       0
   235.2    .045       0   274.3      .1       0     350     .08       0
     380      .1       0
Bank Sta=235.2,274.3
XS Rating Curve= 0 ,0
Exp/Cntr(USF)=0,0
Exp/Cntr=0.3,0.1

Type RM Length L Ch R = 1 ,28239   ,345.1,323.2,296.9
XS GIS Cut Line= 3
2364247.26279239717251.4275748262364699.88621036717330.816741409
2365087.67480865 717398.76133353
#Sta/Elev= 30
       0 2323.13    45.6 2322.97   118.7 2325.41   126.8 2324.65     137 2320.12
   154.3 2320.84   164.7 2316.67   179.6 2313.58     204 2312.82   244.2 2304.43
   274.8 2304.49   338.8 2303.42   382.7 2306.48     407 2306.14   431.4 2302.81
   447.1 2304.11   455.8 2306.54   500.4 2307.03   561.3 2305.29   589.8 2300.62
   626.3 2304.92   642.6 2303.11   654.8 2306.97     671 2318.93   711.6 2353.49
   723.8 2362.24   755.5 2391.66   796.7 2424.04   821.2 2434.91   853.2 2443.28
#Mann= 6 ,-1,0
       0      .1       0      80     .06       0   274.8    .045       0
   338.8      .1       0     380     .08       0  479.53      .1       0
Bank Sta=274.8,338.8
XS Rating Curve= 0 ,0
Exp/Cntr=0.3,0.1

Type RM Length L Ch R = 1 ,27916   ,257.3,267.7,272.5
XS GIS Cut Line= 4
2364001.95967136717621.9529119712364667.64302614717587.137291701
2364793.04497295717499.2213582122365028.62160368717515.014779315
#Sta/Elev= 30
       0 2372.48    66.3 2347.86   146.4 2329.01   230.5 2325.75   269.3 2318.39
   306.6 2318.66   318.7 2316.03   330.7 2316.41   346.7 2323.18   381.9 2321.49
   406.8 2318.58   426.8    2308   450.8 2307.73   462.8 2301.71   490.9 2305.13
     547 2302.96     570 2305.61   666.6 2303.99     677 2301.28   704.8 2299.99
   767.6 2300.05   802.4 2302.44   833.9  2299.1   851.1 2300.69     887 2323.14
   935.1 2347.67     971 2371.13   999.3 2386.74  1019.3  2396.5  1055.8 2409.92
#Mann= 5 ,-1,0
       0      .1       0     320     .06       0     520      .1       0
   704.8    .045       0   767.6      .1       0
Bank Sta=704.8,767.6
XS Rating Curve= 0 ,0
Exp/Cntr(USF)=0,0
Exp/Cntr=0.3,0.1

Type RM Length L Ch R = 1 ,27648   ,269,256.3,251.2
XS GIS Cut Line= 3
2364055.42892725718089.3820938012364640.81976008 717840.31476244
2365069.20852192 717690.66476244
#Sta/Elev= 30
       0 2365.33    13.9 2366.41    48.6 2364.89   126.9 2349.91   144.3 2344.46
   157.3 2338.19   170.3 2329.95   192.1 2320.67   209.5 2316.74   275.2 2312.88
   339.9 2310.89   366.7 2307.57     510 2303.04   539.8 2300.42   577.1  2302.3
   625.9 2301.99   688.6  2298.7   744.9 2301.33   779.6 2300.54   792.3 2298.64
   844.9 2298.16   876.8 2298.55   889.3 2301.73   906.7 2314.96   923.9 2323.25
   957.5 2343.85   995.6 2361.59  1024.4 2370.67  1059.2 2379.56  1089.9 2390.81
#Mann= 7 ,-1,0
       0      .1       0     400     .12       0     420      .1       0
     510     .06       0     610      .1       0   792.3    .045       0
   876.8      .1       0
Bank Sta=792.3,876.8
XS Rating Curve= 0 ,0
Exp/Cntr=0.3,0.1

Type RM Length L Ch R = 1 ,27392   ,236,240.5,243.6
XS GIS Cut Line= 2
2363944.14002125718539.0273399852365076.00186699717928.348390655
#Sta/Elev= 30
       0 2323.72    13.7 2318.67    48.6 2319.68    63.4 2317.26    86.4  2319.3
   122.8 2315.22   145.5 2318.79   186.4 2318.09   204.6 2314.75   243.5 2317.66
   281.8 2317.15   322.7 2336.29   352.7  2344.5   372.7 2345.18   422.7 2332.21
   463.6  2310.9   486.4 2303.11     650  2304.5   695.4  2299.6   763.6 2301.42
     880 2298.46  1034.7 2298.54  1054.5 2296.79    1141 2296.31  1168.1 2295.96
  1170.5 2296.15  1191.1 2298.89    1217 2319.39  1231.8 2329.05  1286.1 2344.47
#Mann= 6 ,-1,0
       0      .1       0     540     .12       0     670     .06       0
     880      .1       0    1141    .045       0  1170.5      .1       0
Bank Sta=1141,1170.5
XS Rating Curve= 0 ,0
Exp/Cntr(USF)=0,0
Exp/Cntr=0.3,0.1

Type RM Length L Ch R = 1 ,27151   ,296.5,288.2,282
XS GIS Cut Line= 3
2363891.43865997718823.2250521222364872.73776008718258.846667061
2365271.76609301718143.858809833
#Sta/Elev= 30
       0 2365.47   116.3  2347.1   188.6 2340.78   208.5 2335.49   242.3 2335.37
   351.5 2327.12   365.4 2325.16   397.2 2312.24   429.3 2309.34   476.1 2308.53
   499.2 2311.27   517.6 2306.47   541.7 2304.31     654 2305.91   758.3 2299.84
   942.4 2300.96  1025.2 2296.38  1082.5 2297.76  1108.3 2294.79  1129.9 2296.65
  1243.8 2296.19  1318.8 2293.69  1345.1 2293.17  1354.7 2294.08  1364.6 2296.55
  1385.4 2310.44    1427 2345.79  1456.1 2374.45  1485.3 2393.64  1547.3 2427.09
#Mann= 5 ,-1,0
       0      .1       0     950     .06       0    1070      .1       0
  1318.8    .045       0  1354.7      .1       0
#XS Ineff= 2 , 0
           943.4 2313.81
Permanent Ineff=
       F       F
Bank Sta=1318.8,1354.7
XS Rating Curve= 0 ,0
Exp/Cntr=0.3,0.1

Type RM Length L Ch R = 1 ,26863   ,213.1,209.5,206.9
XS GIS Cut Line= 2
 2364053.8959972719193.3709607452365324.20823681718368.243675201
#Sta/Elev= 30
       0 2390.51    19.1 2385.13     141 2362.07   212.9 2351.39   250.7 2338.94
   274.6 2337.64   288.9 2332.44   336.6 2324.16   422.5 2315.19   465.4 2302.95
     494  2299.2   632.3 2299.91     720 2297.03   918.4 2296.72   969.7 2294.13
  1023.4 2297.57  1195.2 2297.58  1242.9 2296.51  1257.2 2290.71  1295.3 2293.77
  1314.6 2290.93    1343 2290.46  1375.3  2290.8  1389.7 2293.22  1395.6 2297.02
  1433.6  2333.8    1462 2358.06  1476.3 2366.65  1495.7  2373.1  1514.8 2382.87
#Mann= 6 ,-1,0
       0      .1       0     910     .06       0    1070     .08       0
    1140      .1       0  1314.6    .045       0  1375.3      .1       0
#XS Ineff= 2 , 0
         1024.06 2313.92
Permanent Ineff=
       F       F
Bank Sta=1314.6,1375.3
XS Rating Curve= 0 ,0
Exp/Cntr(USF)=0,0
Exp/Cntr=0.3,0.1
