HEC-RAS study GLADYFK.prj: GLADYFK

--- GLADYFK.g01 (geometry) --- (continued)

Type RM Length L Ch R = 1 ,26654   ,244.1,240.8,239.6
XS GIS Cut Line= 3
2364275.38023165719432.2639093492365087.37609301718806.920287319
2365492.14185545718480.005096561
#Sta/Elev= 30
       0 2374.65    26.2  2366.8    46.4 2357.08    81.8 2355.49   105.4 2345.62
   173.9  2326.1   302.2 2299.79   571.5 2296.38   785.2 2297.05   904.7 2292.97
   975.4 2293.97     995 2297.01  1014.6 2292.97    1067 2290.74  1097.7 2294.59
  1133.9 2295.34  1159.6 2292.25  1185.3 2294.14  1205.9    2289  1221.3 2292.45
  1242.9 2292.83  1265.6 2292.65    1283 2289.35  1344.7 2289.53  1358.7 2293.51
  1376.6 2305.61  1401.3 2327.55  1411.5 2339.85  1428.7 2353.71  1545.2 2433.06
#Mann= 9 ,-1,0
       0      .1       0     310     .08       0     380      .1       0
     430     .12       0     680      .1       0    1020     .06       0
 1054.89      .1       0    1283    .045       0  1344.7      .1       0
#XS Ineff= 2 , 0
          994.91 2350.35
Permanent Ineff=
       F       F
Bank Sta=1283,1344.7
XS Rating Curve= 0 ,0
Exp/Cntr=0.3,0.1

Type RM Length L Ch R = 1 ,26413   ,274.7,279.3,283
XS GIS Cut Line= 2
2364533.62116321719661.5827227762365661.93475368718633.051966841
#Sta/Elev= 30
       0 2375.17   109.7 2345.53   143.1 2333.27   174.8  2315.3     206 2303.67
     250 2296.68   704.3 2292.96   736.9 2296.33   809.9  2295.2   843.7 2296.77
   907.3 2292.04   918.2 2295.56     929 2296.12   950.6 2291.69   999.4 2293.72
  1021.9 2288.39  1037.2 2288.09  1072.4 2291.91  1129.3 2292.18  1210.4 2290.66
  1221.3  2287.4  1267.8 2287.02  1296.1 2287.83  1318.7 2299.39  1348.4 2322.65
  1366.9 2333.04  1394.5 2356.55  1405.3 2362.34    1432 2382.38  1526.8  2440.9
#Mann= 8 ,-1,0
       0      .1       0     240     .08       0     250     .12       0
     830      .1       0     910     .06       0    1050      .1       0
  1221.3    .045       0  1296.1      .1       0
#XS Ineff= 2 , 0
          926.17 2327.26
Permanent Ineff=
       F       F
Bank Sta=1221.3,1296.1
XS Rating Curve= 0 ,0
Exp/Cntr(USF)=0,0
Exp/Cntr=0.3,0.1

Type RM Length L Ch R = 1 ,26134   ,504.5,505.1,505.7
XS GIS Cut Line= 4
2364707.78458423719572.8423524982365309.19915984719278.793406461
2365456.50594676719156.4587635992365844.17499942718884.534658275
#Sta/Elev= 30
       0 2304.22     9.3 2300.63    26.6 2300.25    53.9 2296.22     459 2294.63
   538.3 2290.79   614.9  2290.4   659.4 2291.64   684.1 2294.74   709.6  2290.9
   751.3 2291.36   800.5 2286.27   857.3  2289.3   875.2    2288     909 2290.76
   919.2 2290.15   929.3 2286.03   997.3 2289.91  1064.1 2286.44    1110 2285.82
  1129.3 2286.16  1152.2 2289.78  1159.2 2293.05  1173.1  2304.6    1222 2336.43
  1249.8 2351.22  1265.1 2361.57  1277.6 2366.93  1299.5 2382.25  1334.5 2402.41
#Mann= 9 ,-1,0
       0      .1       0     120     .08       0     170     .12       0
     340      .1       0     390     .12       0     620     .06       0
  789.45      .1       0  1064.1    .045       0  1129.3      .1       0
#XS Ineff= 2 , 0
          683.78 2318.52
Permanent Ineff=
       F       F
Bank Sta=1064.1,1129.3
XS Rating Curve= 0 ,0
Exp/Cntr=0.3,0.1

Type RM Length L Ch R = 1 ,25628   ,506.9,504.7,503.2
XS GIS Cut Line= 3
2365018.70320892720127.975527775 2365713.7328941719588.657816261
2366238.19363137719229.385105324
#Sta/Elev= 30
       0    2388    82.9 2374.72   158.8 2355.04   211.2  2332.5   280.3 2292.22
   447.4 2289.34   462.6 2291.49   493.9 2289.57   558.8 2290.96     574 2287.62
   598.3 2286.92   660.1 2286.57   678.7 2289.29   702.7 2285.41   857.5 2289.12
   887.5 2282.22   911.8 2284.52   940.9  2282.8  1056.6 2286.28  1086.3 2285.94
  1100.9 2281.66  1154.8 2282.48  1171.7 2284.48  1232.7  2281.1  1255.2 2286.04
  1285.1 2311.93  1309.8 2329.31  1388.4  2372.4  1459.2 2419.11  1515.4 2453.02
#Mann= 6 ,-1,0
       0      .1       0     390     .12       0     620     .06       0
     740      .1       0  1100.9    .045       0  1154.8      .1       0
#XS Ineff= 2 , 0
          679.25 2317.76
Permanent Ineff=
       F       F
Bank Sta=1100.9,1154.8
XS Rating Curve= 0 ,0
Exp/Cntr=0.3,0.1

Type RM Length L Ch R = 1 ,25124   ,265.1,259.8,262.1
XS GIS Cut Line= 4
2365431.32275771720517.6193370762366078.89318898719955.409477485
2366470.00935423 719648.18220049     2366592.794      719520.653
#Sta/Elev= 30
       0 2348.46    12.9 2344.34    43.4  2326.8    55.6 2321.87      80 2316.67
   117.7 2302.38   128.3 2301.79   183.7 2288.68     500 2283.59   684.3  2282.4
   721.5  2285.8   818.3 2283.48   920.2 2284.55   968.3 2281.47   990.7 2277.16
  1048.1  2280.3  1072.8 2276.65  1103.4 2276.29  1126.7 2276.73  1133.9 2279.48
  1170.6 2309.71  1201.9 2329.22  1269.1 2364.93  1281.4 2369.16  1375.3 2419.13
  1392.4 2424.27  1429.3 2441.32  1454.8  2449.1  1511.3 2472.74    1532 2478.59
#Mann= 8 ,-1,0
       0      .1       0     350     .12       0     490      .1       0
     500     .12       0     750     .06       0  877.57      .1       0
  1072.8    .045       0  1126.7      .1       0
#XS Ineff= 2 , 0
          775.13 2325.38
Permanent Ineff=
       F       F
Bank Sta=1072.8,1126.7
XS Rating Curve= 0 ,0
Exp/Cntr=0.3,0.1

Type RM Length L Ch R = 1 ,24864   ,334,331.7,329.4
XS GIS Cut Line= 2
2365656.06645423 720644.59891142 2366600.8052145719868.339629453
#Sta/Elev= 30
       0 2344.35    30.9 2326.28    99.1 2296.68   124.4 2289.35   156.6 2285.87
   290.1    2284   312.3 2286.25   351.9 2283.31   417.4 2284.16     443 2282.42
   653.3 2280.27   775.5 2282.13   795.4 2279.73   805.6 2281.12   883.5 2281.14
   914.8 2278.34   926.1 2275.08   947.5 2274.53     989 2275.09   999.3 2279.44
  1019.9 2296.48  1030.4    2303  1051.1 2312.52  1079.6 2329.67  1095.4 2341.37
  1113.7 2352.47  1123.6 2362.99  1184.8 2387.58  1201.2 2399.28  1222.7  2409.1
#Mann= 7 ,-1,0
       0      .1       0     260     .08       0     310      .1       0
     700     .06       0     880      .1       0   926.1    .045       0
     989      .1       0
Bank Sta=926.1,989
XS Rating Curve= 0 ,0
Exp/Cntr(USF)=0,0
Exp/Cntr=0.3,0.1

Type RM Length L Ch R = 1 ,24532   ,387.7,387.5,371.6
XS GIS Cut Line= 2
2366020.34534212720880.9800289512366787.92013948720110.459801755
#Sta/Elev= 30
       0 2337.31    27.9 2324.71    61.8 2315.11   124.4 2313.52   135.5 2311.17
   147.1 2306.29   169.8 2306.17     186 2302.45   203.8 2300.84   277.5 2300.66
     378  2292.2   415.5 2292.39   434.5 2289.09   521.2 2282.28   536.1 2278.19
     553 2276.14   572.2 2277.92   645.9 2276.42   678.6 2279.18   739.4 2276.72
   767.6 2278.09   787.6 2274.77   807.1 2274.45   811.5 2274.36   852.3 2274.42
   910.5 2279.51   950.1 2299.48   967.1 2305.15   995.3  2319.3  1087.6 2358.01
#Mann= 5 ,-1,0
       0      .1       0     560     .06       0     700      .1       0
   807.1    .045       0   852.3      .1       0
Bank Sta=807.1,852.3
XS Rating Curve= 0 ,0
Exp/Cntr(USF)=0,0
Exp/Cntr=0.3,0.1

Type RM Length L Ch R = 1 ,24145   ,260.9,249.2,222.8
XS GIS Cut Line= 3
2366477.43519714721056.1814739582366869.31868437720538.244526042
     2367065.014      720136.074
#Sta/Elev= 30
       0 2341.81    21.2 2331.01      69 2316.03   132.6  2303.6   238.2  2292.5
   255.4 2286.53   276.3 2274.34   299.7  2275.2   354.9 2272.13   375.8 2273.74
   392.9 2272.04   408.9 2274.41   449.5 2273.88   469.5 2276.06   489.5 2273.69
   512.4 2274.94   532.4 2272.56   605.7 2272.99   676.4 2274.64   770.8 2273.02
   788.6 2270.78   833.1 2272.08   859.7 2276.02   873.9 2283.67   904.2 2303.79
   913.1 2306.57   930.9 2317.19   985.1 2335.46  1064.4  2359.2  1096.7 2372.26
#Mann= 5 ,-1,0
       0      .1       0     350     .06       0     510      .1       0
   532.4    .045       0   605.7      .1       0
Bank Sta=532.4,605.7
XS Rating Curve= 0 ,0
Exp/Cntr=0.3,0.1

Type RM Length L Ch R = 1 ,23895   ,265.3,273.8,262.3
XS GIS Cut Line= 4
2366977.29352479721222.3159380122367036.01188511720804.379373381
2367049.82796989 720576.413974492367062.60699515720269.681388379
#Sta/Elev= 30
       0 2333.09    61.7 2293.14   106.2 2273.15   146.6 2267.92     191 2267.29
   207.2 2270.14   243.5 2270.87   259.7 2269.41   271.8 2272.95   287.9 2272.28
   308.1 2274.06   352.6 2272.96     393 2270.06   485.7 2274.79   497.4  2274.2
   515.9 2270.61   570.3 2270.93   605.6 2272.11   657.7 2270.31   673.7 2273.73
   685.7 2273.83   709.6 2272.97   717.7 2271.12   729.7 2272.64   781.8 2272.51
   825.8 2269.29   865.8 2273.23   914.5 2305.65   937.9 2318.03   957.4 2326.37
#Mann= 5 ,-1,0
       0      .1       0     250     .06       0  452.04      .1       0
   515.9    .045       0   570.3      .1       0
Bank Sta=515.9,570.3
XS Rating Curve= 0 ,0
Exp/Cntr(USF)=0,0
Exp/Cntr=0.3,0.1

Type RM Length L Ch R = 1 ,23622   ,161.7,163,163.8
XS GIS Cut Line= 3
2367247.74773646721295.375303384 2367288.1714474720796.357961197
2367295.09114505720378.663303384
#Sta/Elev= 30
       0 2340.64    26.3 2326.12    95.2 2280.12   110.6 2271.47   118.6 2268.62
   154.8 2269.37   186.8 2266.75   198.8 2269.05   214.9 2269.81   232.6 2266.65
     251  2265.6   275.1 2270.78     292 2272.04   411.5 2271.87   463.7 2268.91
   503.8 2271.56   515.8 2268.26   547.8 2267.45   611.8 2272.83   619.8 2272.06
   627.8 2268.57   667.9 2268.59   719.5 2268.35   775.9  2269.7   795.9 2267.95
   803.9 2269.21   811.9 2273.27   835.9 2292.86   867.9 2311.85   918.4 2328.91
#Mann= 5 ,-1,0
       0      .1       0     230     .06       0     320      .1       0
   667.9    .045       0   719.5      .1       0
Bank Sta=667.9,719.5
XS Rating Curve= 0 ,0
Exp/Cntr=0.3,0.1

Type RM Length L Ch R = 1 ,23459   ,303.2,312.9,319.3
XS GIS Cut Line= 3
2367389.78209897721295.4182151582367437.95751608720776.613895645
2367459.85136416720476.789351924
#Sta/Elev= 30
       0 2333.17    14.3 2325.89    30.4 2315.46    50.5 2298.46    70.5 2277.73
    86.6 2266.42   102.7 2264.24   126.8 2265.08   154.9 2268.53     175 2267.23
   211.1 2269.44   243.3 2267.64   263.4 2270.69   283.5 2268.82   303.5 2270.68
   343.7 2267.49   367.8 2269.72     420 2266.39   436.1 2268.46   480.3 2269.64
   563.7 2266.64   576.6 2271.24   628.8  2269.6   642.2 2270.97   683.3 2267.05
   725.7 2266.55   745.1 2266.95   749.1 2268.46   776.7 2287.25   821.7 2312.02
#Mann= 5 ,-1,0
       0      .1       0     230     .06       0     320      .1       0
   683.3    .045       0   725.7      .1       0
Bank Sta=683.3,725.7
XS Rating Curve= 0 ,0
Exp/Cntr(USF)=0,0
Exp/Cntr=0.3,0.1

Type RM Length L Ch R = 1 ,23146   ,148.5,148.2,148
XS GIS Cut Line= 4
2367686.67304457 721303.29500296 2367717.2989091 720753.61807318
2367768.57110554720646.9719427362367768.57091664720513.444586601
#Sta/Elev= 30
       0  2343.2    17.6 2331.93    42.2 2312.13    50.2 2301.73    66.2 2288.17
    82.2 2269.39    98.2 2263.76   134.3 2263.34   206.4 2267.05   222.5 2264.36
   234.9 2264.46   246.5 2267.16   278.5 2267.55   402.7 2265.28   434.8 2268.45
   454.8 2263.42   494.9 2267.37     583 2265.18   627.9 2265.02   639.8 2265.48
   653.1 2268.73   674.7 2266.14   686.7 2266.56     707 2280.68   718.7 2286.94
     747 2307.34   758.7 2313.31   766.7 2319.84   774.7 2321.97   802.4 2334.62
#Mann= 5 ,-1,0
       0      .1       0     130     .06       0     330      .1       0
     583    .045       0   627.9      .1       0
Bank Sta=583,627.9
XS Rating Curve= 0 ,0
Exp/Cntr=0.3,0.1

Type RM Length L Ch R = 1 ,22998   ,447.8,451.7,441.9
XS GIS Cut Line= 4
2367824.21010952721363.7974988472367854.46596032720811.622688294
2367897.26481521720719.998955978 2367901.6763828720544.868096242
#Sta/Elev= 30
       0 2404.37    26.7 2393.65    34.7 2384.21    54.7 2365.57   110.8 2321.52
   138.8 2297.31   142.8 2292.51   150.8  2276.5   154.9 2270.99   166.9 2263.75
   210.9 2262.57     235 2265.94     259 2262.62     279 2262.68   315.1 2267.49
   371.2 2265.77   431.3 2266.43   439.3 2263.99   467.3 2262.14   523.4 2265.91
   580.2 2264.17   628.3 2263.78   639.6 2263.89     657 2267.29     693 2266.16
     705 2263.74     737 2264.34   796.3 2310.28     813 2321.65   829.3 2329.54
#Mann= 5 ,-1,0
       0      .1       0     190     .06       0     290      .1       0
   580.2    .045       0   628.3      .1       0
Bank Sta=580.2,628.3
XS Rating Curve= 0 ,0
Exp/Cntr(USF)=0,0
Exp/Cntr=0.3,0.1

Type RM Length L Ch R = 1 ,22546   ,240.6,235.8,223.1
XS GIS Cut Line= 3
2368072.70329463721346.9024648242368079.44684943721147.224882168
2368277.36488379720425.902834688
#Sta/Elev= 30
       0 2408.83   129.8 2329.27   143.2 2306.83   149.8 2297.68   161.8 2286.28
   173.8  2278.5   185.8 2266.23   189.8 2263.88   210.2 2264.67   218.5 2259.77
   226.8 2259.52   250.9  2259.2   270.4 2260.68   313.9 2263.51   376.1 2261.05
   442.9 2265.42   496.4 2263.74   615.4 2264.71   633.3 2262.31   683.1 2262.78
   699.7 2261.06   720.4 2261.75     739 2264.84     766 2264.66   795.1 2270.01
   807.5 2273.92     849 2293.98   881.9  2306.7   908.3 2314.57   947.8 2323.71
#Mann= 5 ,-1,0
       0      .1       0      80     .06       0   226.8    .045       0
   270.4     .06       0  279.79      .1       0
Bank Sta=226.8,270.4
XS Rating Curve= 0 ,0
Exp/Cntr=0.3,0.1

Type RM Length L Ch R = 1 ,22310   ,188.5,184.8,184.9
XS GIS Cut Line= 3
2368349.22133121721329.2572868942368290.50297089720811.154107598
2368349.22133121720455.389924482
#Sta/Elev= 30
       0  2449.7   116.8 2363.91   128.9 2347.07     149 2333.09   165.1 2315.02
   173.2 2309.31   213.4 2267.21   217.5 2264.45   233.6 2263.98   245.6 2257.78
   253.1 2257.51   268.6 2257.35   285.9 2257.59     306 2260.21   330.2 2258.41
   346.3  2261.7   374.5 2261.95   418.7 2258.15   438.9 2261.93   479.1 2259.05
   547.7 2262.83     568 2260.15   620.7 2263.31   632.9 2260.16   661.3    2260
   684.7 2263.97   746.4 2265.04   762.6 2272.81   778.8 2276.06     882 2287.79
#Mann= 4 ,-1,0
       0      .1       0   253.1    .045       0   285.9     .06       0
     360      .1       0
Bank Sta=253.1,285.9
XS Rating Curve= 0 ,0
Exp/Cntr(USF)=0,0
Exp/Cntr=0.3,0.1

Type RM Length L Ch R = 1 ,22125   ,234.3,238.4,243.6
XS GIS Cut Line= 3
2368571.51639965 721288.317355752368459.60049097720867.289241538
2368424.48545699720454.906770618
#Sta/Elev= 30
       0 2464.92    47.8 2424.22    57.6  2410.8     115 2370.16   127.4 2357.73
   139.4 2350.35   153.1 2338.62   168.8 2321.39   218.5 2284.23     235 2263.95
   257.1 2262.81   268.1 2257.29   275.9 2256.05   284.7 2255.93   321.9 2256.31
   345.4 2260.07   367.5 2259.35   379.9 2256.58   391.1  2260.1   408.9 2261.43
   473.9 2258.34   526.1 2263.93   562.2 2260.95   594.3 2261.83   610.4 2260.22
   738.9 2269.31     775 2275.52   807.1  2290.7   819.1  2294.6   849.5  2298.1
#Mann= 5 ,-1,0
       0      .1       0     230     .06       0   275.9    .045       0
   321.9     .06       0     330      .1       0
Bank Sta=275.9,321.9
XS Rating Curve= 0 ,0
Exp/Cntr=0.3,0.1

Type RM Length L Ch R = 1 ,21887   ,260.9,258,254.7
XS GIS Cut Line= 2
2368753.34181106721215.2745874492368677.35334476720465.751988068
#Sta/Elev= 30
       0 2428.54    14.2 2416.97    42.3 2396.03    54.4  2388.4    74.5 2371.21
   102.6 2348.93     138 2322.65   158.9 2308.46   185.5 2287.38   211.2  2262.5
   231.3 2261.58   239.3  2256.5   251.4 2255.18   267.5 2255.12   309.6 2255.24
   320.6 2255.47   335.8 2257.37   347.9 2255.62     368  2255.4     380 2258.68
   392.1 2257.86   404.2 2259.48   424.3 2260.19   500.6 2260.54     514 2262.08
   633.3 2264.58   645.5 2268.66   685.7 2288.31   717.8 2293.33   753.4 2296.29
#Mann= 5 ,-1,0
       0      .1       0     150     .06       0     240      .1       0
   251.4    .045       0   309.6      .1       0
Bank Sta=251.4,309.6
XS Rating Curve= 0 ,0
Exp/Cntr(USF)=0,0
Exp/Cntr=0.3,0.1

Type RM Length L Ch R = 1 ,21629   ,220.2,225.1,233.7
XS GIS Cut Line= 2
2369037.10535547721162.413316665 2368891.1484474720481.976013281
#Sta/Elev= 30
       0 2406.73    38.9 2385.62    50.4 2378.17    62.5 2373.45      86 2357.37
    95.4 2354.19     169  2308.9   185.4 2297.44   205.8  2280.1   222.2 2260.86
   226.3  2259.4   242.6 2259.53   246.7 2258.18   250.8 2254.93     259 2253.97
   295.8 2253.74     304 2253.91   320.4 2254.84   361.3 2253.99   375.7 2256.46
   399.3 2256.76   426.7 2259.53   451.3 2260.28   467.6 2262.23   479.9 2265.49
   493.6  2265.6   504.5 2268.02   608.1  2277.3     664  2275.3   695.9 2279.81
#Mann= 4 ,-1,0
       0      .1       0     190     .06       0     259    .045       0
     304      .1       0
Bank Sta=259,304
XS Rating Curve= 0 ,0
Exp/Cntr=0.3,0.1

Type RM Length L Ch R = 1 ,21404   ,273.2,271.1,270
XS GIS Cut Line= 2
2369212.72663003721111.6539515892369171.27837569720393.217542967
#Sta/Elev= 30
       0 2367.08    34.5 2356.57    74.6  2340.4   106.7 2326.62   114.7  2322.3
   126.7 2313.46   139.2 2297.35   162.7  2280.2   180.6 2262.45   186.8 2258.41
   206.8 2258.29   226.9 2252.81   234.9 2253.69   246.9 2253.03   274.9    2252
     323 2253.23   351.1 2259.23   363.1 2258.26   391.1 2259.25   427.2 2255.41
   451.2 2255.15   461.3 2258.81   482.5 2273.06   503.3 2284.51   515.3 2288.39
   635.5 2304.46   695.6 2308.67   703.7 2308.38   711.7 2305.96   719.6 2305.64
#Mann= 5 ,-1,0
       0      .1       0     140     .06       0     240      .1       0
   246.9    .045       0     323      .1       0
Bank Sta=246.9,323
XS Rating Curve= 0 ,0
Exp/Cntr(USF)=0,0
Exp/Cntr=0.3,0.1

Type RM Length L Ch R = 1 ,21133   ,239.5,242.9,271.9
XS GIS Cut Line= 3
2369409.80485664721196.043618485 2369476.3914763720886.426334121
      2369408.93      720348.406
#Sta/Elev= 30
       0 2331.04   101.1 2312.97   129.8 2300.64     187 2269.27   203.4 2261.39
   216.5 2257.24     228 2255.41   277.1 2256.36   297.5 2253.65   305.7 2254.27
     330 2249.75   373.2  2250.3   382.4 2249.63   418.7 2250.09   434.9 2253.88
   479.2 2252.66   511.5 2256.16   543.7 2255.56   555.8 2252.99   586.7 2253.97
   597.4 2256.49   622.5 2270.15   636.4 2279.56   647.6  2283.6     713 2294.55
   769.5 2301.41   789.6 2305.76   797.7 2305.22     842 2313.71   858.9 2320.24
#Mann= 7 ,-1,0
       0      .1       0     130     .06       0     140      .1       0
     230     .06       0   326.7      .1       0   373.2    .045       0
   418.7      .1       0
Bank Sta=373.2,418.7
XS Rating Curve= 0 ,0
Exp/Cntr=0.3,0.1

Type RM Length L Ch R = 1 ,20890   ,227.9,253.1,281.6
XS GIS Cut Line= 3
2369506.31843163721194.550460277 2369679.0194914720911.320722262
2369796.45621204720324.137119061
#Sta/Elev= 30
       0 2308.58    20.3 2305.08    48.5 2292.83    63.5 2284.93    85.9  2269.7
   111.1 2255.88   115.9 2254.44   139.1 2254.89   159.5  2253.4     338 2255.07
   350.2  2254.3   362.5 2251.36   427.7 2251.88     440 2249.03   460.3 2248.94
   545.3 2248.97   603.1 2248.98   668.4 2246.94   676.6 2247.39   684.4 2250.46
     697 2266.71     701 2270.08   705.1 2271.95   725.1  2275.4   745.9 2282.34
   782.6 2305.18     852 2352.03   888.8 2369.51     909  2381.2   930.5    2389
#Mann= 5 ,-1,0
       0      .1       0      60     .06       0     250      .1       0
   460.3    .045       0   545.3      .1       0
Bank Sta=460.3,545.3
XS Rating Curve= 0 ,0
Exp/Cntr(USF)=0,0
Exp/Cntr=0.3,0.1

Type RM Length L Ch R = 1 ,20637   ,274.7,285.3,292.5
XS GIS Cut Line= 3
2369540.18523756721298.6750953792369874.81452311 720909.41709597
2370162.31199941720670.619287318
#Sta/Elev= 30
       0 2296.47    54.7 2296.33    85.9  2293.3   116.6 2282.73   154.9 2258.87
   165.5 2254.09     176 2251.69     384 2252.99     405 2254.08   490.9 2252.19
   503.1 2253.43     520 2250.09   530.7 2246.07     540 2245.71   551.4 2244.62
   613.9 2245.97   676.4 2246.25   684.9 2247.73   690.6 2251.17   701.9 2261.03
   712.7 2268.03   733.5 2285.24   758.7 2300.29   775.1 2307.61   789.1  2312.2
   811.5 2317.27   821.2 2318.04   841.1 2324.22   868.7 2340.84   887.1 2347.32
#Mann= 5 ,-1,0
       0      .1       0     150     .06       0     300      .1       0
     540    .045       0   613.9      .1       0
Bank Sta=540,613.9
XS Rating Curve= 0 ,0
Exp/Cntr=0.3,0.1

Type RM Length L Ch R = 1 ,20351   ,189.7,194.8,202.5
XS GIS Cut Line= 2
2369621.72314342721303.3736895232370357.42965802720978.695697164
#Sta/Elev= 30
       0 2283.98    33.3 2278.85    46.4  2274.7    64.9 2267.58    94.5 2252.23
   103.2 2249.98   133.8 2251.44   161.3  2250.2     265 2250.64   369.9 2252.89
   439.9 2249.94   444.3 2249.02     453 2244.13   467.6 2243.71   482.8 2242.94
   524.8 2243.22   544.8  2244.6   549.6 2246.61   566.7 2262.76   592.9  2284.2
   610.2  2295.7   622.4 2301.71   634.5 2305.53   645.4 2312.06     689  2349.8
   698.2 2355.08   713.4 2359.67   741.6 2371.87   789.2 2401.46   804.2 2408.35
#Mann= 5 ,-1,0
       0      .1       0      80     .06       0     130      .1       0
   467.6    .045       0   524.8      .1       0
Bank Sta=467.6,524.8
XS Rating Curve= 0 ,0
Exp/Cntr(USF)=0,0
Exp/Cntr=0.3,0.1

Type RM Length L Ch R = 1 ,20156   ,227.5,235.6,244.7
XS GIS Cut Line= 2
2369532.65923697      721407.7882370365.73200236721246.600475712
#Sta/Elev= 30
       0    2287    40.2 2280.48   117.7 2274.25     134 2271.85   158.4 2264.95
     191 2250.28     210 2249.61   227.7 2250.84   292.8 2249.03   337.7 2250.86
     391 2250.04   419.1 2251.16   451.7 2249.03   504.7 2250.06   537.3 2248.23
   557.7 2241.47   561.7 2241.38   606.6 2241.07   614.7 2241.16   626.9 2241.55
   636.8  2244.2   651.4 2252.73   671.7 2269.25     688 2279.91   696.2 2283.65
   720.6 2298.55   776.7 2329.47   818.4 2348.73   838.8 2360.16   848.5 2364.15
#Mann= 7 ,-1,0
       0      .1       0     110     .06       0     200      .1       0
     210     .06       0     310      .1       0   561.7    .045       0
   614.7      .1       0
Bank Sta=561.7,614.7
XS Rating Curve= 0 ,0
Exp/Cntr=0.3,0.1

Type RM Length L Ch R = 1 ,19921   ,262.6,269.1,274.2
XS GIS Cut Line= 2
2369569.91282549721458.8046433112370374.69976399721565.879300366
#Sta/Elev= 30
       0 2278.85    66.8 2269.36      83 2268.23   103.2 2261.19   123.3 2250.21
   127.4 2249.54   151.6 2250.38   179.8 2247.59   191.9 2249.45   232.3 2247.44
   268.6 2250.42   357.4 2249.81   417.9 2247.49   462.3 2248.23   494.6  2246.2
   525.8  2239.4   555.1 2239.26   579.3 2239.53   591.4 2240.12   599.5 2243.93
   631.8 2270.47   643.9 2278.24     660 2292.64   679.4 2307.73   712.8  2331.7
   720.6 2335.83   749.2 2355.22     773 2368.93   789.2  2376.7   811.9 2391.37
#Mann= 5 ,-1,0
       0      .1       0      70     .06       0     170      .1       0
   525.8    .045       0   579.3      .1       0
#XS Ineff= 2 , 0
          266.82 2264.32
Permanent Ineff=
       F       F
Bank Sta=525.8,579.3
XS Rating Curve= 0 ,0
Exp/Cntr(USF)=0,0
Exp/Cntr=0.3,0.1

Type RM Length L Ch R = 1 ,19652   ,214.9,218.2,219.5
XS GIS Cut Line= 2
2369467.85204621721588.4958566362370226.38304917721853.040381515
#Sta/Elev= 30
       0 2289.18    25.9  2277.6    46.9 2270.95    85.1 2260.75      95 2253.95
     102 2251.24     123 2251.79   140.1 2249.12   152.8 2249.46   245.8 2246.38
   288.4 2248.39   355.7 2246.11   415.1 2248.92   445.2  2247.6   555.3 2246.99
   563.8 2245.72   575.6 2238.84   581.9 2237.82   597.3 2237.38   645.9 2238.09
     658  2238.4   666.7 2241.04   673.9 2245.07   695.1 2260.58   699.3 2265.79
     712 2287.14   720.5 2298.69   724.7 2302.89     764 2335.49   803.3 2361.63
#Mann= 4 ,-1,0
       0     .06       0     180      .1       0   581.9    .045       0
   645.9      .1       0
#XS Ineff= 2 , 0
          377.05 2267.24
Permanent Ineff=
       F       F
Bank Sta=581.9,645.9
XS Rating Curve= 0 ,0
Exp/Cntr=0.3,0.1

Type RM Length L Ch R = 1 ,19433   ,283.8,283.1,283
XS GIS Cut Line= 2
2369369.57959616721735.1263389362370236.53891618722108.160628028
#Sta/Elev= 30
       0 2298.63    59.4 2267.31    76.6 2253.66    96.3  2252.8   113.1 2247.48
   211.8  2247.9   233.6 2245.57   285.9 2245.73   307.6 2243.31   325.1 2246.22
   338.1 2244.77   346.8 2246.94   486.2 2244.19   560.7 2246.01     582 2243.72
   599.4 2236.73   609.4 2236.42     656 2236.29   673.3 2236.53   686.5  2237.4
   708.3 2247.03   747.5 2274.05     791 2307.94   808.4 2319.93   845.2 2339.82
   856.3 2344.65   874.3 2350.34   886.8 2356.58   934.7 2385.16   943.8 2389.47
#Mann= 3 ,-1,0
       0      .1       0   609.4    .045       0   673.3      .1       0
#XS Ineff= 2 , 0
          326.17 2267.26
Permanent Ineff=
       F       F
Bank Sta=609.4,673.3
XS Rating Curve= 0 ,0
Exp/Cntr(USF)=0,0
Exp/Cntr=0.3,0.1

Type RM Length L Ch R = 1 ,19150   ,248.6,245.9,242.3
XS GIS Cut Line= 2
 2369246.0222984721989.709482264 2370077.2652984722347.436575008
#Sta/Elev= 30
       0  2309.6    34.7 2292.12      53 2285.14    67.7 2278.08    89.4 2263.01
   102.5 2262.78   111.2  2261.3   124.3 2251.82   141.7 2245.98   294.1 2244.14
   307.2 2245.46   424.7 2245.71   437.8 2242.53   446.5 2244.08   498.8 2244.33
     551 2241.41   568.5 2236.82   581.5 2238.74   598.9 2235.22   620.7 2234.86
   694.7 2235.35   707.6 2236.45   725.2 2243.63   744.1 2254.64   764.4 2269.43
   790.5 2284.27   820.2 2296.91   851.5 2313.19   868.9 2323.82   904.9 2348.92
#Mann= 5 ,-1,0
       0      .1       0     110     .06       0     210      .1       0
   598.9    .045       0   694.7      .1       0
#XS Ineff= 2 , 0
          446.58 2259.75
Permanent Ineff=
       F       F
Bank Sta=598.9,694.7
XS Rating Curve= 0 ,0
Exp/Cntr=0.3,0.1

Type RM Length L Ch R = 1 ,18904   ,256.1,255.3,255.6
XS GIS Cut Line= 2
2369203.78657879722280.861687794 2370077.6539412722588.269574175
#Sta/Elev= 30
       0 2298.62    42.8 2275.34    72.1 2261.36      81 2254.85    85.2 2253.31
   106.4 2253.15   132.3 2244.78   148.8 2243.15   229.4 2241.94   259.1 2241.94
   267.5 2243.31   279.7 2241.86   318.4 2242.85   361.3 2240.51     416 2240.73
   437.2 2242.17     505 2237.78     522 2233.34   530.4 2233.32   615.3 2233.84
   631.1  2238.1   661.9 2240.75   670.4 2244.35   693.8 2260.24   713.1 2277.32
   767.9 2316.01   776.4 2320.39   814.5 2344.99   863.2 2379.11   926.4 2419.29
#Mann= 5 ,-1,0
       0      .1       0      40     .06       0     150      .1       0
     522    .045       0   615.3      .1       0
Bank Sta=522,615.3
XS Rating Curve= 0 ,0
Exp/Cntr(USF)=0,0
Exp/Cntr=0.3,0.1

Type RM Length L Ch R = 1 ,18649   ,276.7,275.7,275.1
XS GIS Cut Line= 2
2369177.51024113722552.1421112922369979.11271554722815.923039843
#Sta/Elev= 30
       0 2280.36    37.8 2261.51    53.3 2250.75    57.5 2249.43    74.4 2249.68
    85.3 2244.48    95.4 2242.12   120.7 2241.42   158.6 2243.01   204.9 2239.05
   259.6 2237.94   289.2 2239.28   338.8  2238.5   373.6  2240.4   394.4 2237.34
   430.7 2235.47   448.2 2232.74   474.4 2232.06   525.7 2232.07   541.8 2232.75
   562.9 2237.62   575.5 2241.91     605 2257.64   647.1 2284.55   677.8 2306.66
   722.9 2332.88   745.5 2350.06   798.7 2383.25   807.1 2389.67   843.9 2411.64
#Mann= 5 ,-1,0
       0      .1       0      70     .06       0     180      .1       0
   448.2    .045       0   525.7      .1       0
Bank Sta=448.2,525.7
XS Rating Curve= 0 ,0
Exp/Cntr=0.3,0.1

Type RM Length L Ch R = 1 ,18373   ,224.2,223,222.5
XS GIS Cut Line= 2
2369120.66755448722832.8215781552369900.23461183723073.037008616
#Sta/Elev= 30
       0 2266.21    25.5 2253.84    49.7  2254.4    62.3 2250.33   104.1 2245.85
   120.9 2245.83   141.8 2243.03     192 2239.78   234.7 2239.05   263.2 2234.25
     305 2233.81   355.3 2235.68   376.2 2232.24   401.3 2234.27     418 2231.43
   428.6 2231.32   449.5 2231.08   490.2 2231.42   501.8 2231.65   526.9 2235.43
   543.6 2242.58   577.1 2262.31   593.8 2274.86   626.1  2294.9   670.2 2325.81
   702.7 2346.51   727.8 2365.43   761.4 2388.09   782.2 2401.09   815.7 2419.18
#Mann= 5 ,-1,0
       0      .1       0      30     .06       0     130      .1       0
   428.6    .045       0   490.2      .1       0
Bank Sta=428.6,490.2
XS Rating Curve= 0 ,0
Exp/Cntr(USF)=0,0
Exp/Cntr=0.3,0.1

Type RM Length L Ch R = 1 ,18150   ,291.1,286.5,281.4
XS GIS Cut Line= 2
2369091.03578584723063.7271720362369820.23907434723273.867743718
#Sta/Elev= 30
       0 2255.64     9.5 2253.92    24.7 2244.02    34.4 2241.26   171.9    2238
   180.2 2236.34   196.8 2236.45   207.5 2234.58   241.2 2235.61   259.3 2232.66
   288.4 2232.32   318.8 2234.55   325.9 2233.84   334.2 2229.35   342.5 2228.83
   363.3 2230.39     430 2229.69   457.7 2231.17   484.1 2234.48   504.9 2233.97
   525.9 2241.45     559 2257.48     587 2274.94   625.8 2297.17   650.6 2313.61
   658.9 2320.84   708.9 2352.14     738 2367.14   750.5 2374.66   758.9 2378.07
#Mann= 4 ,-1,0
       0     .06       0      60      .1       0   363.3    .045       0
     430      .1       0
Bank Sta=363.3,430
XS Rating Curve= 0 ,0
Exp/Cntr=0.3,0.1

Type RM Length L Ch R = 1 ,17864   ,204.9,203,201.2
XS GIS Cut Line= 2
2369070.81152174723417.4968711642369764.26361345723483.216187045
#Sta/Elev= 30
       0  2272.9    17.4 2269.53    61.6 2258.37    89.8    2256    97.8 2253.66
   112.8 2245.91   121.9 2242.61   186.2 2242.73   194.2 2240.45   210.2 2239.54
   224.8 2236.57   250.5 2236.34   282.6 2228.42   301.9 2227.83   353.3 2227.49
     375 2230.16   395.1 2231.33   403.2 2230.56   419.2 2232.15   455.4 2230.22
   467.4 2227.53   495.6 2231.87   503.6 2232.07   527.7 2238.97   543.8 2246.23
   555.8 2254.33   577.2 2266.41     596 2280.08   672.1 2329.13   696.6 2342.13
#Mann= 5 ,-1,0
       0      .1       0      80     .06       0     270      .1       0
   301.9    .045       0   353.3      .1       0
Bank Sta=301.9,353.3
XS Rating Curve= 0 ,0
Exp/Cntr(USF)=0,0
Exp/Cntr=0.3,0.1

Type RM Length L Ch R = 1 ,17661   ,255.2,258,259
XS GIS Cut Line= 3
 2369107.0107016723643.7778431862369520.54334407      723654.331
2369742.77749911723640.035728495
#Sta/Elev= 30
       0  2265.9   101.2  2257.4   129.2 2256.16   145.2 2254.25   157.2 2248.25
   177.2 2247.35   189.2 2239.75   197.2 2237.15   209.2 2230.66   224.9 2229.95
   237.2 2227.29   248.3 2226.86   293.3  2226.7   305.3 2227.75   317.3 2228.26
   337.3 2226.69   349.3 2232.02   377.5 2231.93   417.3 2229.43   429.3 2229.63
   440.8 2227.51   445.4 2225.48   453.4 2224.54   473.4 2229.88   505.5 2240.27
   537.6 2255.95   561.3 2268.85   577.6 2279.02   593.7 2291.33   636.4 2318.14
#Mann= 5 ,-1,0
       0      .1       0      40     .06       0     240      .1       0
   248.3    .045       0   305.3      .1       0
Bank Sta=248.3,305.3
XS Rating Curve= 0 ,0
Exp/Cntr=0.3,0.1

Type RM Length L Ch R = 1 ,17403   ,151.2,149.5,146
XS GIS Cut Line= 3
2368957.84896999723864.9008850172369437.95791614 723906.34913936
2369700.46352698723826.906651868
#Sta/Elev= 30
       0 2307.67    22.4 2303.88    62.6 2295.18   126.8 2277.79   142.8 2274.38
   224.2 2264.34   243.2 2259.42   255.3 2252.41   259.3 2251.08   275.3  2250.5
   279.4 2248.94   319.5 2225.92   331.3 2225.68   387.8  2225.6   411.9 2225.89
   431.9 2229.54   472.1 2228.66   484.2  2229.5   534.4  2229.2   587.3 2227.93
   609.7 2228.97     643 2223.73   647.2 2223.91   668.1 2229.69   677.1 2234.96
   693.2 2241.32   705.7 2249.81   718.2 2253.65   739.1 2262.98   756.2 2274.98
#Mann= 5 ,-1,0
       0      .1       0     290     .06       0   331.3    .045       0
   387.8     .06       0     390      .1       0
Bank Sta=331.3,387.8
XS Rating Curve= 0 ,0
Exp/Cntr(USF)=0,0
Exp/Cntr=0.3,0.1

Type RM Length L Ch R = 1 ,17253   ,288.5,283.4,278.5
XS GIS Cut Line= 3
2369057.90942614724053.4125620362369617.20166679724021.096920946
2369739.36351172723967.563889089
#Sta/Elev= 30
       0 2263.92    34.3 2258.19    98.4 2257.41   114.5 2255.74   138.5 2250.51
   154.5 2250.09   178.6 2237.63   186.6 2231.98   194.6 2225.03   206.9 2224.03
   252.4 2223.78   278.6  2226.5   294.8 2224.42   306.8 2227.43   314.8  2228.2
   358.9  2226.5   370.9 2227.61   398.9 2225.95     419 2228.09     463 2227.76
   495.1 2226.34   527.1 2227.59   547.2 2225.23   563.5 2221.05   571.5 2223.09
   576.6 2225.49   589.7 2227.12   611.5 2236.71   659.7 2262.44   693.6 2283.95
#Mann= 5 ,-1,0
       0      .1       0      90     .06       0     190      .1       0
   206.9    .045       0   252.4      .1       0
Bank Sta=206.9,252.4
XS Rating Curve= 0 ,0
Exp/Cntr=0.3,0.1

Type RM Length L Ch R = 1 ,16970   ,272.1,255.3,217.2
XS GIS Cut Line= 3
2369116.16930092724387.626982841 2369629.2676035724231.895529209
2369803.00832365724094.837988533
#Sta/Elev= 30
       0 2273.77    66.9 2266.97   142.1 2260.94   146.3 2258.99   167.2  2242.5
   183.9 2240.51   200.8  2226.8   204.8 2224.73   213.6 2223.54   234.1 2223.31
   306.6 2223.57   317.7 2222.51     347 2226.59   457.3 2225.06   482.5 2223.52
   497.4 2224.86   535.1 2224.22   557.3 2225.54   590.9 2223.39   597.2 2220.69
   605.7 2219.69   622.8 2223.84   641.8 2222.99   646.9 2223.97     657 2231.43
   668.4 2241.61   692.8 2255.86   733.5 2275.85   743.7 2279.78   757.5 2287.61
#Mann= 5 ,-1,0
       0     .06       0      30      .1       0     140     .06       0
   234.1    .045       0   306.6      .1       0
Bank Sta=234.1,306.6
XS Rating Curve= 0 ,0
Exp/Cntr(USF)=0,0
Exp/Cntr=0.3,0.1

Type RM Length L Ch R = 1 ,16715   ,343.7,354,369.3
XS GIS Cut Line= 3
2369394.90881306724776.840406532 2369610.6589759724376.096021919
 2369831.7163324724120.498453468
#Sta/Elev= 30
       0 2249.41    40.5 2247.38    74.5 2239.77      95 2244.15   112.4 2243.18
   126.8 2240.58     172 2242.54   190.4 2238.37   213.1 2238.49   276.7 2233.45
   299.4 2225.13   326.7 2224.21   340.3 2221.03   358.5 2220.44   402.3 2220.22
   426.6 2222.48   449.4 2221.32   469.6 2223.82   522.4 2222.91   602.9  2224.5
   614.2 2222.59   622.9  2223.6   634.1 2220.07   640.9 2219.56   659.9 2221.48
     671 2225.55   693.6 2242.35   712.8 2252.27   744.6 2265.95   793.1 2290.18
#Mann= 5 ,-1,0
       0      .1       0     100     .06       0     300      .1       0
   358.5    .045       0   402.3      .1       0
Bank Sta=358.5,402.3
XS Rating Curve= 0 ,0
Exp/Cntr=0.3,0.1

Type RM Length L Ch R = 1 ,16361   ,246.1,236.5,229.3
XS GIS Cut Line= 2
2369446.42035175724810.087701217 2370030.7354599724340.468337486
#Sta/Elev= 30
       0 2245.92    22.8 2244.01    38.2 2237.91    43.3 2237.08    70.2 2238.57
    87.2 2236.71   122.8 2235.29   161.1 2235.62   192.1 2233.27   202.4 2230.79
   303.5 2225.37   326.2 2225.35   346.2 2221.81   376.9 2223.87   417.3 2224.66
   469.2 2223.98   494.9 2225.92   522.6 2224.67   531.4 2223.15   550.6 2223.13
   576.92217.958   592.4 2217.42   627.32217.525   633.5 2219.48   647.7 2228.67
   665.5 2237.84   689.9 2256.92   718.9 2263.71   742.1 2276.24   749.6 2278.96
#Mann= 4 ,-1,0
       0     .06       0     120      .1       0   576.9    .045       0
   627.3      .1       0
Bank Sta=576.9,627.3
XS Rating Curve= 0 ,0
Exp/Cntr(USF)=0,0
Exp/Cntr=0.3,0.1

Type RM Length L Ch R = 1 ,16124   ,218.2,219.1,219.6
XS GIS Cut Line= 2
2369680.15947012725186.0405048662370155.40659347724491.711448922
#Sta/Elev= 30
       0 2274.69    35.4 2247.53    56.7 2229.18    83.4 2223.08   102.8 2222.67
   158.9 2224.84   176.2 2220.74   204.6 2221.64   219.2 2217.67   233.7 2219.88
   294.1 2222.92   335.5 2221.92   354.1  2218.9   403.5  2222.9     510 2222.81
   563.3 2221.37   602.1 2222.09   616.1 2219.88   623.2 2220.81   644.5 2220.32
   658.6 2217.53     670 2216.96   674.8 2216.91   729.5 2217.56   737.8 2217.84
   747.5 2221.51   771.9 2242.79   781.5 2249.79   814.4 2269.31   841.4 2281.92
#Mann= 5 ,-1,0
       0      .1       0     100     .06       0     220      .1       0
     670    .045       0   729.5      .1       0
#XS Ineff= 2 , 0
          150.37 2239.45
Permanent Ineff=
       F       F
Bank Sta=670,729.5
XS Rating Curve= 0 ,0
Exp/Cntr=0.3,0.1

Type RM Length L Ch R = 1 ,15905   ,243,229.4,220.7
XS GIS Cut Line= 2
2369838.21127386725256.6520963722370370.76435082 724579.06328781
#Sta/Elev= 30
       0 2273.18    14.6 2265.73      42 2247.85      55 2238.59    70.6 2225.08
    86.5 2223.44   106.4 2216.33     152 2220.31   184.4 2221.61   223.3 2221.35
   251.7 2219.53   294.4  2219.5   319.8 2220.76   370.7 2217.63   436.9 2221.75
   508.1 2220.66   533.5 2217.93   553.4 2218.82   564.1 2216.91   579.3 2216.12
   650.5 2216.53   669.9 2217.12   686.2  2219.6   691.2  2221.1   702.3 2227.32
   728.2 2247.35   761.6 2277.64   792.9 2302.75   823.5 2321.61   861.8 2340.81
#Mann= 5 ,-1,0
       0      .1       0      60     .06       0     190      .1       0
   579.3    .045       0   650.5      .1       0
Bank Sta=579.3,650.5
XS Rating Curve= 0 ,0
Exp/Cntr(USF)=0,0
Exp/Cntr=0.3,0.1

Type RM Length L Ch R = 1 ,15676   ,283.1,264.7,256.6
XS GIS Cut Line= 3
2370221.72483044725351.547466296 2370379.8635337724984.292635859
2370487.83263968724708.802013552
#Sta/Elev= 30
       0 2269.75    28.7 2253.49    49.3 2243.03    76.7 2231.57      94 2226.16
   115.8 2223.29   128.9 2219.12   163.7 2218.21   181.1 2214.72   220.3 2217.56
   272.6 2218.04   289.8 2216.39   299.5 2217.46   320.5 2215.49   420.4 2215.21
   445.7 2215.62   467.6 2218.17   479.7 2217.44   506.3 2217.92   510.6 2216.97
   516.7 2213.86   521.3 2213.06   522.9 2213.09   543.2 2213.37   562.2 2217.74
   572.3 2222.59   640.2 2263.67   656.7 2274.08     671 2284.76   695.7 2300.06
#Mann= 5 ,-1,0
       0      .1       0      50     .06       0     260      .1       0
   522.9    .045       0   543.2      .1       0
Bank Sta=522.9,543.2
XS Rating Curve= 0 ,0
Exp/Cntr=0.3,0.1

Type RM Length L Ch R = 1 ,15411   ,286.1,275.5,271.5
XS GIS Cut Line= 2
2370836.37741959725384.7766142222370609.75908897 724725.31727211
#Sta/Elev= 30
       0 2288.82      25  2274.9    46.1 2264.29    54.6 2261.14    86.8 2242.22
   111.4 2226.72   126.5 2219.12   134.9  2215.9   144.6 2214.81   160.3  2215.9
   177.2  2214.9   207.6 2215.65   220.2 2213.58   232.2 2214.68   257.6 2214.77
   291.4 2212.45   380.2 2212.63   437.4 2211.61   456.6 2211.97   497.2 2211.65
   515.6 2213.55   560.2 2215.86   583.3 2215.69   587.5  2216.5   594.8 2220.18
   617.1  2235.2   638.2 2251.12   646.7  2255.5   667.8 2269.97   697.3 2287.38
#Mann= 5 ,-1,0
       0      .1       0      90     .06       0     190      .1       0
   456.6    .045       0   497.2      .1       0
Bank Sta=456.6,497.2
XS Rating Curve= 0 ,0
Exp/Cntr(USF)=0,0
Exp/Cntr=0.3,0.1

Type RM Length L Ch R = 1 ,15135   ,259.4,260.1,259
XS GIS Cut Line= 3
2371277.06948749 725165.719402712370978.45136924724863.113010455
2370767.45725817724617.000067407
#Sta/Elev= 30
       0 2307.19    35.4 2287.56    46.3 2283.78    73.8 2266.57      83 2264.07
     100 2254.55   146.9 2233.44   167.9 2215.29   187.7 2209.88   196.2    2210
   219.9 2214.34   253.6 2212.64   298.6 2214.71   320.2 2212.94   349.2 2213.58
   388.5    2209   490.9 2212.24   521.7 2209.28   575.2 2208.92   582.3  2209.6
   612.5 2212.85   633.2 2210.31     656 2219.25   674.9 2239.28   686.8 2248.31
   697.6 2258.99   706.9 2264.25     728 2281.89   742.1  2289.1   749.3 2294.94
#Mann= 5 ,-1,0
       0      .1       0     100     .06       0     240      .1       0
   521.7    .045       0   582.3      .1       0
Bank Sta=521.7,582.3
XS Rating Curve= 0 ,0
Exp/Cntr=0.3,0.1

Type RM Length L Ch R = 1 ,14875   ,312.6,299,270.6
XS GIS Cut Line= 3
2371400.65706285724940.6046862022371022.20445071724521.360774549
2370820.51413645724453.375275362
#Sta/Elev= 30
       0 2285.33    24.6 2271.61    79.2 2235.38   101.6 2221.85   113.2 2215.06
   127.4 2208.78   179.8  2211.6     235 2211.38   245.5 2210.88   257.4 2207.68
   275.3 2207.12   317.1 2209.47     335 2209.11   352.9 2210.72   399.3 2211.44
   419.5 2207.41   433.2 2207.14   472.3 2207.49   516.5 2210.38     588 2208.31
   604.9 2206.66   629.7 2211.29   642.9 2211.46   655.6 2215.62     664 2222.25
     677  2238.3   692.8 2249.25   731.6 2268.43   769.5 2283.73   777.6 2287.95
#Mann= 5 ,-1,0
       0      .1       0      40     .06       0     290      .1       0
   433.2    .045       0   472.3      .1       0
Bank Sta=433.2,472.3
XS Rating Curve= 0 ,0
Exp/Cntr(USF)=0,0
Exp/Cntr=0.3,0.1

Type RM Length L Ch R = 1 ,14576   ,232.2,229.6,227.3
XS GIS Cut Line= 3
2371656.75510598724497.6763679632371486.51216574724447.648788047
2370762.30147012724327.092646456
#Sta/Elev= 30
       0 2332.19    21.5 2325.89    54.8  2311.4    75.6 2294.78    96.5 2281.12
     109 2277.53     159 2251.28   179.8  2242.3   204.1 2236.33   220.4 2234.07
   273.1 2229.48   289.3 2215.08   301.5 2214.01   313.7 2205.55   334.6 2204.84
   350.1 2204.56   393.7 2204.92   552.9 2209.24   573.1 2207.24   609.6 2207.85
   646.1 2205.95   702.9 2210.44   755.6 2209.29     780 2217.78   796.2 2226.73
   808.3 2229.66   824.3  2240.6   848.9 2251.24   865.1 2261.33   911.6 2281.02
#Mann= 4 ,-1,0
       0      .1       0  267.44     .06       0   334.6    .045       0
   393.7      .1       0
Bank Sta=334.6,393.7
XS Rating Curve= 0 ,0
Exp/Cntr=0.3,0.1

Type RM Length L Ch R = 1 ,14347   ,200.4,198.9,197.6
XS GIS Cut Line= 3
2371550.72974191724215.7061227952371173.21904135724172.465231451
2370810.62971235724104.479732264
#Sta/Elev= 30
       0 2305.06    42.8 2274.26    58.9 2264.52    83.1 2252.85   119.3 2237.75
   159.9 2230.67   163.6 2229.13   175.7 2217.24   179.7 2215.08   195.8 2212.36
   203.9  2204.6   227.4 2202.95   235.8 2202.85   268.3 2203.09   280.4  2203.6
   288.4 2206.19   312.6 2207.37   413.6 2208.62   454.3 2207.58   462.9 2204.91
     495 2208.81   531.6 2209.47   564.2  2208.3   580.5 2204.33     613 2204.52
   625.2 2207.61   649.6  2207.8   681.8 2224.83   694.4  2229.9   748.9 2238.07
#Mann= 5 ,-1,0
       0      .1       0      50     .06       0     150      .1       0
   227.4    .045       0   268.3      .1       0
Bank Sta=227.4,268.3
XS Rating Curve= 0 ,0
Exp/Cntr(USF)=0,0
Exp/Cntr=0.3,0.1

Type RM Length L Ch R = 1 ,14148   ,263.5,260.5,256.6
XS GIS Cut Line= 3
2371614.48395083724011.7994283182371137.87099823723976.257142773
2370734.81790344723955.373095379
#Sta/Elev= 30
       0 2337.78    74.5 2299.36   114.6 2274.19   138.7 2255.83   150.7 2248.37
   191.2 2213.06   198.9 2210.25   210.9 2209.66   222.9 2204.67     255 2202.22
   315.2 2202.11   335.2  2202.4   351.7 2204.93   367.3 2204.59   383.4 2201.74
   407.4 2206.01   443.5 2206.13   459.6 2202.76   471.6 2206.27   551.7 2207.98
   599.8 2207.13   615.8 2202.97   638.6 2202.61   655.9 2206.84   683.9 2206.99
   703.9 2213.91     720 2217.02   796.1 2226.53   836.1 2226.11   881.5 2234.02
#Mann= 4 ,-1,0
       0      .1       0     210     .06       0     255    .045       0
   315.2      .1       0
Bank Sta=255,315.2
XS Rating Curve= 0 ,0
Exp/Cntr=0.3,0.1

Type RM Length L Ch R = 1 ,13887   ,227.1,229.2,230.2
XS GIS Cut Line= 2
2371518.18250019723731.8184774622370704.78123282723741.144334689
#Sta/Elev= 30
       0 2329.32      46 2294.18      78 2267.31     118 2238.34     146 2211.83
     154 2207.38     162  2206.9     174 2200.39   189.2  2200.1   219.2 2199.93
     286 2202.61     338 2198.35     354 2202.15     386 2204.66   430.5 2204.74
   450.2 2200.76   462.1 2200.91     478 2204.38     498 2204.34     514 2200.55
     522 2200.17     550 2201.75     562 2204.75     594 2203.43     614 2205.26
   682.1 2206.39   722.1 2211.83   778.1 2214.97   797.8 2222.66   813.5 2225.78
#Mann= 5 ,-1,0
       0      .1       0     120     .06       0   189.2    .045       0
   219.2     .06       0     220      .1       0
Bank Sta=189.2,219.2
XS Rating Curve= 0 ,0
Exp/Cntr(USF)=0,0
Exp/Cntr=0.3,0.1

Type RM Length L Ch R = 1 ,13658   ,277.3,275.6,274.8
XS GIS Cut Line= 4
2371488.10552547723519.4245716822371188.91834193723499.242018291
2370883.00408735723466.5297096222370743.68020663723385.600652194
#Sta/Elev= 30
       0 2296.05      40 2268.86    88.1 2238.96   100.2 2229.96     111 2218.09
   128.2 2204.02   140.2 2203.68   148.3 2199.49   160.3 2198.64   200.4  2198.9
   216.4  2199.4   224.4 2202.23   232.5 2202.21     369 2199.54   385.1 2197.54
   413.3 2199.59   425.3 2202.16   437.4 2198.72   453.5 2197.92   469.6 2202.44
   505.8 2201.22   525.9 2204.62     550 2203.45   590.3 2205.32   610.8 2210.44
   639.8  2211.8   657.1 2210.71   670.9 2213.87   705.8 2225.92   768.6 2253.99
#Mann= 4 ,-1,0
       0      .1       0      90     .06       0   160.3    .045       0
   200.4      .1       0
Bank Sta=160.3,200.4
XS Rating Curve= 0 ,0
Exp/Cntr=0.3,0.1

Type RM Length L Ch R = 1 ,13383   ,204.8,212.7,230
XS GIS Cut Line= 3
2371628.97368405723366.7111670142371437.60709374723233.258150092
2370908.83098896 723230.74016864
#Sta/Elev= 30
       0 2304.38    56.3 2274.37    59.5 2272.11    72.6 2258.36   103.4 2242.03
   142.5 2215.71   163.5 2204.96   170.5 2202.49     196 2197.59   210.7 2199.57
   234.8 2198.78   262.7 2200.88   322.7 2202.14   338.7 2196.82   350.3 2196.59
   370.2 2196.62   375.3 2196.81   386.7 2200.55   390.7 2200.78   421.9 2196.17
   466.7 2196.52   490.7 2198.92   514.7 2195.88   526.7  2196.3   554.7 2199.76
   570.7 2200.06   618.7 2206.75   684.7 2209.24   724.5 2215.86   762.1 2228.19
#Mann= 5 ,-1,0
       0      .1       0     160     .06       0   273.3      .1       0
   350.3    .045       0   370.2      .1       0
Bank Sta=350.3,370.2
XS Rating Curve= 0 ,0
Exp/Cntr(USF)=0,0
Exp/Cntr=0.3,0.1

Type RM Length L Ch R = 1 ,13170   ,308.6,333.4,361
XS GIS Cut Line= 3
2371694.04366588723294.9680947882371443.57957286 723076.96409597
2371011.19333471 722932.40566647
#Sta/Elev= 30
       0 2280.04    63.7  2249.2      88 2234.66   145.7  2204.6   161.1 2198.51
   177.5 2197.79   225.2  2201.3   249.3 2198.82   262.3 2195.69   297.5 2199.22
   348.3 2197.57   407.3 2199.47   424.2 2196.85   453.7 2197.05   466.4  2194.9
     479 2194.96   538.1  2194.7   563.4 2195.76   567.6 2197.65   580.3 2199.13
   644.3 2194.56   660.4 2196.97   668.8 2203.16   685.7 2219.92   697.2  2229.1
     711 2236.95   723.4 2241.87   736.3  2250.5   753.2  2258.1     788 2278.42
#Mann= 5 ,-1,0
       0      .1       0     240     .06       0  372.05      .1       0
     479    .045       0   538.1      .1       0
Bank Sta=479,538.1
XS Rating Curve= 0 ,0
Exp/Cntr=0.3,0.1

Type RM Length L Ch R = 1 ,12837   ,199.7,198.9,198.4
XS GIS Cut Line= 3
 2371740.3901026723186.5351126282371529.80056243722924.504536306
 2371471.0476619722639.133305151
#Sta/Elev= 30
       0 2243.99    27.4 2229.19    47.9  2216.4    58.2 2211.91    78.7 2199.89
    83.6 2198.01      89 2197.16   106.4 2197.05   145.4 2198.67   191.6 2198.41
   237.3  2196.3   255.8 2194.22   289.1 2198.36   328.3 2198.82   347.7 2196.99
   372.2 2196.09   376.3 2195.45   384.6 2191.89   396.7 2191.25     409 2191.15
   437.6 2191.63   449.8 2192.03     458 2194.57   474.3 2205.42   498.8 2224.62
   535.6 2250.17   592.8 2281.89   601.1 2287.84   614.7 2295.52   627.5 2305.05
#Mann= 5 ,-1,0
       0      .1       0      70     .06       0     220      .1       0
   396.7    .045       0   437.6      .1       0
Bank Sta=396.7,437.6
XS Rating Curve= 0 ,0
Exp/Cntr(USF)=0,0
Exp/Cntr=0.3,0.1

Type RM Length L Ch R = 1 ,12638   ,290.6,295,298.3
XS GIS Cut Line= 3
2371860.85980033723189.3783011382371733.25519968722929.951432087
     2371668.679722626.098980379
#Sta/Elev= 30
       0 2269.74    18.1 2260.24    54.4 2236.08    67.1 2229.38    98.3 2208.88
   120.6 2197.17   129.1 2195.91   156.2 2195.64   187.4 2198.36     210 2197.16
   224.8 2198.73   260.6 2198.61   275.6 2194.56   302.2 2192.45   314.4 2195.66
   330.8 2196.71     339 2195.38   351.2 2191.47   367.6 2190.41   408.7 2190.34
   416.7 2190.44     433 2190.61   437.1 2191.15   441.2 2193.27   465.7 2212.95
   494.4 2230.57   514.8 2245.39     568 2278.08   580.7 2284.42   599.7 2295.82
#Mann= 5 ,-1,0
       0      .1       0     170     .06       0     280      .1       0
   367.6    .045       0   416.7      .1       0
Bank Sta=367.6,416.7
XS Rating Curve= 0 ,0
Exp/Cntr=0.3,0.1

Type RM Length L Ch R = 1 ,12343   ,331.9,332.6,333
XS GIS Cut Line= 2
2372026.09309036723152.4213230452371991.97930077722593.808018622
#Sta/Elev= 30
       0 2264.26    23.3    2250    48.4 2236.26    99.4 2206.28   111.4 2201.21
   127.5 2196.54   139.5 2194.38   155.5 2194.13   195.6 2195.45   219.7 2194.64
   231.9 2196.37   243.7 2196.85   259.7 2194.24   271.7 2194.31   287.8 2189.03
     307 2188.78   331.9 2188.75   347.9 2188.79   375.9  2189.4     388 2197.22
     400  2203.4     416    2215     424 2219.76     441 2232.57   452.1 2239.24
   472.1 2253.34   484.1  2263.6   495.9 2271.67   528.2  2296.2   559.7  2317.1
#Mann= 4 ,-1,0
       0      .1       0     210     .06       0     307    .045       0
   347.9      .1       0
Bank Sta=307,347.9
XS Rating Curve= 0 ,0
Exp/Cntr(USF)=0,0
Exp/Cntr=0.3,0.1

Type RM Length L Ch R = 1 ,12010   ,127.5,127.7,127.9
XS GIS Cut Line= 2
2372343.10113488723164.2074248182372335.19663553722636.857763046
#Sta/Elev= 30
       0 2285.71      23 2268.32      35 2260.32      55 2245.27    77.3 2229.77
     103 2209.62     115 2203.06     123 2199.93     127 2199.13     135 2195.68
     163    2194   186.9 2196.27   231.1 2196.28   263.1 2190.27   275.1 2189.65
   285.7 2187.87   300.2 2187.78   354.9 2187.78   377.8 2187.75   387.1 2188.51
   399.1 2194.94   415.8 2204.99   435.1 2218.86     455 2229.04   471.2 2239.01
   482.8 2246.99   499.1 2254.52   511.1  2261.5   523.1 2269.91   527.4 2271.73
#Mann= 5 ,-1,0
       0      .1       0     130     .06       0     220      .1       0
   300.2    .045       0   354.9      .1       0
Bank Sta=300.2,354.9
XS Rating Curve= 0 ,0
Exp/Cntr=0.3,0.1
